HEC-RAS study Chauga River.prj: Chauga River Limited Detail Study

--- Chauga River.g01 (geometry) --- (continued)

Type RM Length L Ch R = 1,121500,395,395,395
BEGIN DESCRIPTION:
Chauga River 243.0
END DESCRIPTION:
XS GIS Cut Line= 3
      1336835.57      1082172.12      1336317.51      1082082.82
      1335419.78      1082157.06
#Sta/Elev= 30
  4474.3 1327.72  4491.8 1322.95  4499.0 1330.13  4510.2 1332.31  4540.6 1331.23
  4628.8 1368.95  4648.9 1371.18  4678.7 1367.16  4753.0 1344.30  4776.2 1332.84
  4837.3 1280.32  4900.3 1241.60  4949.9 1234.16  4964.0 1221.83  4969.9 1226.06
  4975.4 1221.34  4975.9 1220.34  5024.6 1221.34  5034.0 1221.83  5034.7 1226.68
  5041.0 1230.55  5463.5 1233.81  5537.1 1239.47  5582.3 1238.22  5598.7 1242.68
  5598.9 1246.34  5601.3 1241.38  5612.3 1248.02  5713.7 1281.60  5900.8 1302.19
#Mann=3,-1,0
  4474.3    0.15       0  4975.4    0.05       0  5024.6    0.15       0
Bank Sta=4975.4,5024.6
XS Rating Curve= 0
Exp/Cntr=0.3,0.1

Type RM Length L Ch R = 1,121105,523,523,523
BEGIN DESCRIPTION:
Chauga River 242.0
END DESCRIPTION:
XS GIS Cut Line= 3
      1337148.96      1081772.68      1336308.52      1081692.04
      1335675.05      1081675.00
#Sta/Elev= 30
  4155.7 1441.99  4257.1 1400.33  4305.8 1367.26  4370.3 1334.17  4398.5 1311.22
  4452.7 1278.82  4534.5 1268.07  4557.1 1258.80  4558.1 1254.64  4563.1 1258.36
  4692.3 1238.71  4864.6 1234.29  4913.8 1224.67  4940.9 1228.48  4975.2 1220.91
  4975.7 1219.91  5024.8 1220.91  5039.0 1227.83  5119.6 1227.55  5132.1 1235.48
  5350.9 1236.85  5401.3 1254.61  5409.9 1262.95  5443.8 1277.51  5489.2 1291.94
  5498.0 1299.42  5533.0 1300.73  5563.5 1309.39  5600.3 1309.31  5633.7 1319.42
#Mann=3,-1,0
  4155.7    0.15       0  4975.2    0.05       0  5024.8    0.15       0
Bank Sta=4975.2,5024.8
XS Rating Curve= 0
Exp/Cntr=0.3,0.1

Type RM Length L Ch R = 1,120582,582,582,582
BEGIN DESCRIPTION:
Chauga River 241.0
END DESCRIPTION:
XS GIS Cut Line= 3
      1336675.95      1080986.42      1336137.48      1081206.22
      1335775.19      1081356.96
#Sta/Elev= 30
  4418.4 1409.22  4443.3 1394.56  4466.2 1390.70  4472.0 1381.49  4501.0 1373.85
  4510.0 1365.51  4567.2 1348.98  4594.6 1324.97  4668.5 1289.16  4708.0 1262.76
  4772.2 1241.72  4780.9 1237.13  4781.3 1232.32  4783.5 1239.61  4785.3 1240.22
  4798.9 1233.44  4824.7 1229.41  4954.8 1227.66  4975.2 1218.80  4975.7 1217.80
  5024.8 1218.80  5030.1 1222.30  5030.8 1218.80  5032.1 1223.52  5050.4 1231.04
  5065.9 1233.29  5217.0 1232.19  5272.8 1256.38  5348.9 1303.97  5392.4 1309.36
#Mann=3,-1,0
  4418.4    0.15       0  4975.2    0.05       0  5024.8    0.15       0
Bank Sta=4975.2,5024.8
XS Rating Curve= 0
Exp/Cntr=0.3,0.1

Type RM Length L Ch R = 1,120000,609,609,609
BEGIN DESCRIPTION:
Chauga River 240.0
END DESCRIPTION:
XS GIS Cut Line= 3
      1335962.00      1080421.26      1335842.72      1080811.65
      1335742.08      1081439.53
#Sta/Elev= 30
  4591.8 1395.54  4625.4 1381.76  4646.6 1363.85  4659.2 1359.27  4698.4 1357.42
  4728.2 1348.71  4736.5 1351.98  4763.8 1335.63  4828.0 1323.29  4837.0 1314.22
  4884.9 1303.77  4889.9 1295.00  4902.1 1288.90  4915.0 1269.05  4929.3 1260.59
  4946.0 1257.18  4949.7 1238.48  4951.0 1245.33  4951.9 1222.98  4957.5 1234.62
  4975.2 1216.38  4975.7 1215.38  5024.8 1216.38  5033.5 1224.64  5159.0 1230.10
  5265.0 1248.80  5376.6 1257.58  5390.3 1260.16  5425.9 1278.12  5635.9 1320.99
#Mann=3,-1,0
  4591.8    0.15       0  4975.2    0.05       0  5024.8    0.15       0
Bank Sta=4975.2,5024.8
XS Rating Curve= 0
Exp/Cntr=0.3,0.1

Type RM Length L Ch R = 1,119391,475,475,475
BEGIN DESCRIPTION:
Chauga River 239.0
END DESCRIPTION:
XS GIS Cut Line= 3
      1335251.05      1080430.30      1335255.87      1080962.18
      1335371.43      1081351.28
#Sta/Elev= 30
  4468.1 1381.15  4518.9 1362.34  4544.9 1360.52  4581.0 1332.16  4593.5 1315.02
  4604.9 1304.86  4654.2 1279.22  4691.0 1255.68  4718.9 1243.10  4801.6 1229.51
  4866.9 1225.27  4935.0 1226.23  4947.6 1221.36  4950.3 1224.71  4961.9 1221.21
  4964.8 1213.97  4965.7 1216.81  4975.0 1213.97  4975.5 1212.97  5025.0 1213.97
  5031.4 1214.43  5046.7 1224.16  5092.0 1228.66  5148.0 1229.65  5250.7 1241.75
  5286.9 1238.14  5312.9 1246.22  5327.3 1246.42  5343.7 1254.69  5405.9 1266.81
#Mann=3,-1,0
  4468.1    0.15       0  4975.0    0.05       0  5025.0    0.15       0
Bank Sta=4975,5025
XS Rating Curve= 0
Exp/Cntr=0.3,0.1

Type RM Length L Ch R = 1,118916,522,522,522
BEGIN DESCRIPTION:
Chauga River 238.0
END DESCRIPTION:
XS GIS Cut Line= 3
      1335016.34      1080363.71      1334792.91      1081049.85
      1334693.75      1081403.31
#Sta/Elev= 30
  4278.4 1277.89  4308.2 1256.25  4326.0 1251.21  4362.7 1253.46  4386.0 1259.84
  4476.0 1245.45  4526.8 1232.66  4722.8 1223.76  4798.9 1225.47  4825.9 1219.72
  4950.0 1222.97  4966.4 1213.04  4975.0 1213.04  4975.5 1212.04  5025.0 1213.04
  5033.6 1219.01  5035.9 1213.04  5039.6 1226.40  5074.3 1256.48  5120.7 1266.65
  5146.1 1285.39  5156.5 1288.00  5165.9 1297.37  5191.8 1303.34  5206.2 1317.77
  5293.9 1339.21  5294.2 1336.02  5301.7 1335.36  5324.5 1342.69  5367.1 1339.73
#Mann=3,-1,0
  4278.4    0.15       0  4975.0    0.05       0  5025.0    0.15       0
Bank Sta=4975,5025
XS Rating Curve= 0
Exp/Cntr=0.3,0.1

Type RM Length L Ch R = 1,118394,493,493,493
BEGIN DESCRIPTION:
Chauga River 237.0
END DESCRIPTION:
XS GIS Cut Line= 3
      1334913.67      1080219.42      1334346.70      1080802.66
      1333970.75      1081147.28
#Sta/Elev= 30
  4186.6 1380.37  4276.9 1318.02  4285.2 1302.01  4321.2 1276.00  4391.7 1242.32
  4434.2 1230.95  4506.9 1225.26  4632.9 1228.73  4685.4 1225.03  4719.7 1217.89
  4739.8 1223.93  4895.2 1226.65  4927.8 1219.47  4948.9 1220.93  4954.0 1213.04
  4959.6 1223.57  4975.0 1213.04  4975.5 1212.04  5025.0 1213.04  5025.6 1216.12
  5035.3 1213.04  5045.7 1224.13  5109.1 1237.75  5243.7 1296.08  5344.4 1329.00
  5346.1 1324.52  5349.6 1330.15  5399.9 1347.20  5444.5 1359.36  5510.0 1363.66
#Mann=3,-1,0
  4186.6    0.15       0  4975.0    0.05       0  5025.0    0.15       0
Bank Sta=4975,5025
XS Rating Curve= 0
Exp/Cntr=0.3,0.1

Type RM Length L Ch R = 1,117901,401,401,401
BEGIN DESCRIPTION:
Chauga River 236.0
END DESCRIPTION:
XS GIS Cut Line= 3
      1334455.74      1080089.92      1334241.41      1080330.23
      1333925.02      1080774.97
#Sta/Elev= 30
  4678.0 1338.55  4707.6 1330.75  4814.4 1284.02  4846.8 1266.08  4854.4 1259.42
  4866.8 1255.81  4872.1 1251.33  4878.2 1249.62  4892.8 1239.99  4904.2 1230.33
  4929.0 1223.28  4930.7 1216.86  4948.9 1210.70  4957.4 1213.27  4964.8 1210.33
  4975.0 1210.33  4975.5 1209.33  5025.0 1210.33  5028.1 1219.97  5082.2 1219.60
  5097.9 1217.06  5168.7 1219.21  5212.1 1228.88  5231.4 1239.09  5245.9 1241.41
  5326.7 1280.36  5359.7 1294.35  5394.8 1305.50  5435.2 1313.89  5545.8 1323.63
#Mann=3,-1,0
  4678.0    0.15       0  4975.0    0.05       0  5025.0    0.15       0
Bank Sta=4975,5025
XS Rating Curve= 0
Exp/Cntr=0.3,0.1

Type RM Length L Ch R = 1,117500,500,500,500
BEGIN DESCRIPTION:
Chauga River 235.0
END DESCRIPTION:
XS GIS Cut Line= 3
      1334356.37      1080036.87      1333919.72      1080245.87
      1333446.54      1080521.91
#Sta/Elev= 30
  4515.9 1335.27  4616.6 1315.69  4728.9 1278.68  4730.5 1279.23  4731.1 1283.02
  4737.3 1277.59  4753.4 1271.37  4775.8 1267.59  4818.6 1274.34  4836.2 1273.83
  4902.7 1257.16  4911.0 1254.21  4970.9 1217.60  4975.0 1209.51  4975.5 1208.51
  5025.0 1209.51  5054.8 1210.33  5076.6 1217.81  5097.6 1229.25  5114.7 1246.10
  5156.4 1274.11  5159.5 1282.04  5168.3 1280.98  5185.6 1291.83  5213.2 1303.69
  5436.8 1351.74  5466.1 1355.58  5486.7 1362.68  5505.4 1363.68  5547.8 1376.46
#Mann=3,-1,0
  4515.9    0.15       0  4975.0    0.05       0  5025.0    0.15       0
Bank Sta=4975,5025
XS Rating Curve= 0
Exp/Cntr=0.3,0.1

Type RM Length L Ch R = 1,117000,500,500,500
BEGIN DESCRIPTION:
Chauga River 234.0
END DESCRIPTION:
XS GIS Cut Line= 3
      1334244.93      1079693.45      1333879.79      1079767.11
      1333455.59      1079913.37
#Sta/Elev= 30
  4627.5 1343.55  4674.5 1319.34  4718.3 1293.54  4742.4 1275.87  4803.2 1263.92
  4818.3 1255.27  4840.2 1255.13  4858.3 1248.40  4908.4 1225.32  4920.7 1211.17
  4926.0 1208.67  4926.7 1203.16  4936.2 1209.18  4950.4 1203.83  4951.6 1201.82
  4952.6 1194.77  4967.9 1213.80  4973.0 1206.17  4975.0 1194.77  4975.5 1193.77
  5025.0 1194.77  5038.6 1205.81  5064.3 1209.05  5139.5 1204.54  5153.8 1209.98
  5219.2 1212.64  5250.8 1221.87  5320.6 1257.30  5424.0 1323.59  5448.7 1328.49
#Mann=3,-1,0
  4627.5    0.15       0  4975.0    0.05       0  5025.0    0.15       0
Bank Sta=4975,5025
XS Rating Curve= 0
Exp/Cntr=0.3,0.1

Type RM Length L Ch R = 1,116500,500,500,500
BEGIN DESCRIPTION:
Chauga River 233.0
END DESCRIPTION:
XS GIS Cut Line= 3
      1333916.52      1079300.03      1333535.70      1079416.75
      1333320.07      1079553.06
#Sta/Elev= 30
  4601.7 1400.66  4662.7 1373.25  4709.0 1359.28  4780.9 1331.54  4804.2 1316.49
  4825.8 1307.51  4877.7 1278.18  4878.5 1274.74  4879.6 1237.11  4890.9 1239.88
  4895.2 1236.42  4904.6 1237.93  4918.7 1248.92  4919.8 1239.00  4938.3 1216.22
  4949.5 1212.54  4958.9 1223.07  4974.1 1206.06  4974.4 1191.91  4974.9 1190.91
  5025.6 1191.91  5034.8 1195.40  5035.6 1211.42  5036.1 1207.64  5042.9 1191.95
  5097.6 1231.28  5186.9 1284.48  5223.3 1296.05  5237.4 1296.22  5255.1 1289.42
#Mann=3,-1,0
  4601.7    0.15       0  4974.4    0.05       0  5025.6    0.15       0
Bank Sta=4974.4,5025.6
XS Rating Curve= 0
Exp/Cntr=0.3,0.1

Type RM Length L Ch R = 1,116000,500,500,500
BEGIN DESCRIPTION:
Chauga River 232.0
END DESCRIPTION:
XS GIS Cut Line= 3
      1333606.25      1078815.01      1333188.36      1079062.15
      1332829.02      1079312.07
#Sta/Elev= 30
  4514.5 1462.46  4558.4 1450.87  4617.7 1421.70  4707.0 1364.26  4834.6 1294.73
  4915.5 1241.81  4928.6 1239.85  4952.2 1210.95  4957.2 1199.31  4961.1 1203.71
  4973.2 1199.96  4973.6 1187.58  4974.4 1187.58  4974.9 1186.58  5025.6 1187.58
  5029.6 1188.11  5032.7 1206.29  5035.5 1188.39  5041.6 1188.46  5111.1 1242.67
  5133.0 1244.76  5223.1 1305.08  5258.2 1319.96  5295.1 1322.13  5296.9 1317.35
  5325.2 1308.47  5338.5 1324.74  5353.2 1306.61  5357.2 1297.12  5437.7 1270.76
#Mann=3,-1,0
  4514.5    0.15       0  4974.4    0.05       0  5025.6    0.15       0
Bank Sta=4974.4,5025.6
XS Rating Curve= 0
Exp/Cntr=0.3,0.1

Type RM Length L Ch R = 1,115500,500,500,500
BEGIN DESCRIPTION:
Chauga River 231.0
END DESCRIPTION:
XS GIS Cut Line= 3
      1333509.81      1078435.45      1332994.08      1078631.41
      1332624.14      1078851.18
#Sta/Elev= 30
  4448.3 1418.12  4577.9 1338.82  4596.9 1315.68  4613.3 1311.05  4677.3 1265.37
  4704.8 1263.48  4738.6 1242.13  4777.1 1236.83  4877.8 1178.75  4910.3 1189.75
  4920.6 1170.88  4974.4 1165.38  4974.9 1164.38  5025.6 1165.38  5050.7 1169.56
  5070.1 1190.76  5071.3 1208.48  5092.5 1213.43  5130.9 1251.45  5133.7 1246.80
  5161.8 1267.08  5170.1 1284.30  5175.4 1275.90  5260.8 1321.90  5301.9 1353.20
  5324.3 1361.30  5326.1 1355.30  5345.0 1350.01  5360.3 1361.74  5430.3 1330.97
#Mann=3,-1,0
  4448.3    0.15       0  4974.4    0.05       0  5025.6    0.15       0
Bank Sta=4974.4,5025.6
XS Rating Curve= 0
Exp/Cntr=0.3,0.1

Type RM Length L Ch R = 1,115000,500,500,500
BEGIN DESCRIPTION:
Chauga River 230.0
END DESCRIPTION:
XS GIS Cut Line= 3
      1333091.08      1077842.01      1332840.37      1078178.73
      1332509.69      1078607.15
#Sta/Elev= 30
  4580.2 1348.43  4607.1 1347.48  4613.3 1353.50  4726.3 1310.89  4819.7 1253.86
  4870.9 1230.86  4883.2 1218.35  4906.9 1177.27  4924.7 1174.73  4925.0 1161.44
  4929.0 1172.12  4938.9 1168.28  4953.4 1176.63  4974.4 1155.57  4974.9 1154.57
  5025.6 1155.57  5042.6 1166.42  5088.5 1174.80  5163.1 1172.54  5249.7 1186.78
  5328.2 1211.79  5336.0 1226.39  5347.9 1220.41  5354.1 1228.66  5372.7 1226.35
  5384.4 1257.16  5393.1 1262.33  5417.6 1246.80  5463.1 1284.33  5541.2 1312.02
#Mann=3,-1,0
  4580.2    0.15       0  4974.4    0.05       0  5025.6    0.15       0
Bank Sta=4974.4,5025.6
XS Rating Curve= 0
Exp/Cntr=0.3,0.1

Type RM Length L Ch R = 1,114500,500,500,500
BEGIN DESCRIPTION:
Chauga River 229.0
END DESCRIPTION:
XS GIS Cut Line= 3
      1332741.63      1077811.87      1332357.86      1078062.57
      1331856.02      1078474.58
#Sta/Elev= 30
  4541.6 1251.45  4601.2 1269.60  4636.6 1269.24  4805.5 1219.65  4847.6 1198.33
  4862.5 1174.29  4877.3 1170.44  4881.9 1158.66  4890.3 1177.27  4899.2 1171.11
  4902.1 1151.51  4908.6 1169.75  4923.8 1149.03  4927.0 1156.76  4938.1 1150.23
  4974.4 1148.42  4974.9 1147.42  5025.6 1148.42  5067.5 1154.55  5092.0 1177.57
  5159.6 1203.34  5234.5 1219.57  5271.3 1212.45  5325.3 1182.74  5426.0 1230.20
  5471.8 1240.84  5590.6 1285.34  5594.7 1297.31  5603.4 1289.75  5649.3 1304.26
#Mann=3,-1,0
  4541.6    0.15       0  4974.4    0.05       0  5025.6    0.15       0
Bank Sta=4974.4,5025.6
XS Rating Curve= 0
Exp/Cntr=0.3,0.1

Type RM Length L Ch R = 1,114000,500,500,500
BEGIN DESCRIPTION:
Chauga River 228.0
END DESCRIPTION:
XS GIS Cut Line= 3
      1332886.22      1077486.52      1332404.04      1077580.21
      1332118.11      1077599.78
#Sta/Elev= 30
  4508.8 1409.19  4526.9 1404.47  4552.1 1387.41  4561.5 1387.81  4613.2 1344.96
  4637.9 1339.56  4653.1 1324.35  4679.6 1309.04  4694.0 1296.48  4703.6 1295.23
  4714.4 1286.64  4778.3 1258.01  4814.8 1233.50  4834.2 1215.52  4896.9 1185.35
  4898.2 1187.76  4936.9 1155.84  4955.8 1152.10  4959.8 1146.23  4974.4 1146.23
  4974.9 1145.23  5025.6 1146.23  5040.3 1165.95  5061.0 1185.67  5095.7 1204.85
  5131.2 1232.00  5137.4 1240.99  5216.3 1267.23  5246.9 1266.92  5286.6 1250.11
#Mann=3,-1,0
  4508.8    0.15       0  4974.4    0.05       0  5025.6    0.15       0
Bank Sta=4974.4,5025.6
XS Rating Curve= 0
Exp/Cntr=0.3,0.1

Type RM Length L Ch R = 1,113500,500,500,500
BEGIN DESCRIPTION:
Chauga River 227.0
END DESCRIPTION:
XS GIS Cut Line= 3
      1332271.70      1076888.24      1332140.67      1077210.42
      1332027.70      1077602.78
#Sta/Elev= 30
  4652.2 1288.13  4706.2 1281.42  4740.8 1282.57  4805.4 1248.21  4829.2 1228.68
  4855.6 1217.18  4899.9 1181.47  4924.3 1166.36  4927.1 1168.49  4936.9 1145.44
  4940.5 1148.44  4974.4 1141.68  4974.9 1140.68  5025.6 1141.68  5036.4 1147.50
  5050.9 1146.93  5061.9 1154.68  5128.6 1161.36  5137.3 1174.34  5143.8 1174.51
  5145.3 1179.55  5195.7 1186.52  5237.3 1200.78  5259.6 1200.57  5296.9 1211.72
  5301.5 1205.50  5307.7 1211.42  5312.0 1210.37  5378.8 1242.67  5408.3 1249.31
#Mann=3,-1,0
  4652.2    0.15       0  4974.4    0.05       0  5025.6    0.15       0
Bank Sta=4974.4,5025.6
XS Rating Curve= 0
Exp/Cntr=0.3,0.1

Type RM Length L Ch R = 1,113000,500,500,500
BEGIN DESCRIPTION:
Chauga River 226.0
END DESCRIPTION:
XS GIS Cut Line= 3
      1331813.80      1076557.49      1331654.43      1077111.63
      1331449.28      1077575.71
#Sta/Elev= 30
  4423.4 1299.41  4492.9 1283.23  4513.1 1265.98  4573.1 1232.57  4626.6 1210.64
  4721.8 1151.98  4735.3 1156.16  4802.0 1146.02  4934.9 1145.35  4974.4 1136.62
  4974.9 1135.62  5025.6 1136.62  5028.4 1143.64  5038.9 1146.22  5048.1 1159.31
  5068.4 1162.59  5172.5 1154.62  5174.1 1167.25  5227.5 1182.80  5276.2 1213.37
  5319.5 1256.69  5342.7 1265.37  5353.1 1259.41  5363.6 1273.17  5380.8 1274.96
  5415.0 1261.35  5495.4 1219.87  5497.0 1209.14  5502.1 1226.96  5507.4 1227.09
#Mann=3,-1,0
  4423.4    0.15       0  4974.4    0.05       0  5025.6    0.15       0
Bank Sta=4974.4,5025.6
XS Rating Curve= 0
Exp/Cntr=0.3,0.1

Type RM Length L Ch R = 1,112500,500,500,500
BEGIN DESCRIPTION:
Chauga River 225.0
END DESCRIPTION:
XS GIS Cut Line= 3
      1331298.68      1076569.48      1331229.36      1076864.96
      1331093.82      1077346.76
#Sta/Elev= 30
  4696.5 1283.40  4721.0 1277.14  4748.7 1263.27  4817.3 1211.68  4842.2 1200.25
  4881.2 1168.69  4921.7 1148.72  4944.5 1145.58  4974.4 1134.57  4974.9 1133.57
  5025.6 1134.57  5033.1 1134.57  5044.1 1144.61  5049.9 1140.03  5115.1 1142.49
  5132.2 1149.42  5218.2 1145.60  5245.9 1149.23  5255.6 1152.46  5257.9 1158.51
  5258.3 1165.01  5259.6 1158.47  5271.8 1159.02  5332.3 1188.52  5351.0 1203.87
  5394.0 1218.62  5397.6 1225.41  5422.4 1244.15  5443.3 1243.70  5500.5 1256.49
#Mann=3,-1,0
  4696.5    0.15       0  4974.4    0.05       0  5025.6    0.15       0
Bank Sta=4974.4,5025.6
XS Rating Curve= 0
Exp/Cntr=0.3,0.1

Type RM Length L Ch R = 1,112000,500,500,500
BEGIN DESCRIPTION:
Chauga River 224.0
END DESCRIPTION:
XS GIS Cut Line= 3
      1331123.90      1076515.31      1330830.74      1076636.70
      1330470.27      1076798.45
#Sta/Elev= 30
  4682.7 1310.55  4742.9 1292.88  4764.0 1279.62  4793.7 1270.50  4823.3 1245.19
  4857.0 1226.08  4927.7 1160.41  4940.6 1156.36  4941.8 1151.27  4949.8 1142.18
  4952.2 1143.55  4963.3 1132.80  4964.3 1138.42  4973.3 1136.14  4974.0 1132.80
  4974.5 1131.80  5026.0 1132.80  5035.9 1132.80  5041.2 1147.87  5064.4 1144.00
  5085.6 1160.04  5115.0 1171.63  5178.9 1185.61  5210.2 1197.32  5216.7 1205.99
  5254.4 1200.25  5287.2 1218.78  5344.9 1231.03  5380.3 1245.16  5395.1 1242.83
#Mann=3,-1,0
  4682.7    0.15       0  4974.0    0.05       0  5026.0    0.15       0
Bank Sta=4974,5026
XS Rating Curve= 0
Exp/Cntr=0.3,0.1

Type RM Length L Ch R = 1,111500,594,594,594
BEGIN DESCRIPTION:
Chauga River 223.0
END DESCRIPTION:
XS GIS Cut Line= 3
      1330789.55      1076104.39      1330483.83      1076277.04
      1330102.71      1076538.18
#Sta/Elev= 30
  4648.9 1269.84  4696.1 1261.51  4711.4 1244.18  4756.0 1224.58  4763.0 1231.22
  4791.3 1225.42  4877.7 1187.67  4932.0 1174.76  4941.8 1151.03  4956.1 1150.26
  4962.3 1132.55  4974.0 1127.50  4974.5 1126.50  5026.0 1127.50  5036.0 1127.50
  5038.5 1139.76  5039.5 1133.82  5050.9 1138.24  5083.5 1163.75  5091.4 1161.25
  5122.9 1184.46  5271.8 1245.22  5365.9 1291.37  5409.6 1305.76  5416.0 1302.49
  5417.4 1310.11  5425.8 1301.82  5437.8 1300.40  5441.2 1308.22  5462.0 1297.93
#Mann=3,-1,0
  4648.9    0.15       0  4974.0    0.05       0  5026.0    0.15       0
Bank Sta=4974,5026
XS Rating Curve= 0
Exp/Cntr=0.3,0.1

Type RM Length L Ch R = 1,110906,569,569,569
BEGIN DESCRIPTION:
Chauga River 222.0
END DESCRIPTION:
XS GIS Cut Line= 3
      1330554.58      1075715.78      1330076.28      1075844.83
      1329683.96      1076007.99
#Sta/Elev= 30
  4504.6 1228.17  4521.6 1216.25  4544.4 1228.49  4585.4 1230.17  4592.8 1226.26
  4649.5 1232.00  4700.2 1223.43  4801.6 1197.06  4810.1 1191.56  4822.9 1169.11
  4847.8 1175.96  4901.4 1146.81  4943.3 1149.09  4955.3 1129.66  4956.0 1142.50
  4958.6 1141.95  4968.3 1137.40  4974.0 1125.60  4974.5 1124.60  5026.0 1125.60
  5046.2 1134.45  5047.0 1125.60  5057.5 1143.22  5081.1 1134.66  5090.6 1169.29
  5150.3 1193.05  5200.8 1224.28  5275.9 1251.85  5319.2 1262.97  5424.9 1270.57
#Mann=3,-1,0
  4504.6    0.15       0  4974.0    0.05       0  5026.0    0.15       0
Bank Sta=4974,5026
XS Rating Curve= 0
Exp/Cntr=0.3,0.1

Type RM Length L Ch R = 1,110337,582,582,582
BEGIN DESCRIPTION:
Chauga River 221.0
END DESCRIPTION:
XS GIS Cut Line= 3
      1330374.96      1075225.01      1329887.01      1075320.45
      1329388.79      1075515.13
#Sta/Elev= 30
  4502.8 1307.68  4569.9 1300.69  4652.5 1288.10  4683.0 1286.01  4703.8 1278.53
  4758.1 1256.85  4787.4 1242.21  4825.4 1229.90  4842.3 1219.54  4858.7 1205.17
  4869.7 1198.09  4883.9 1175.62  4896.7 1183.93  4909.3 1174.46  4928.0 1152.25
  4937.7 1143.13  4973.6 1129.85  4974.0 1125.73  4974.5 1124.73  5026.0 1125.73
  5030.5 1134.37  5085.1 1142.65  5135.5 1180.05  5207.3 1221.30  5244.7 1237.53
  5282.1 1245.81  5329.7 1252.99  5407.2 1273.50  5456.6 1272.98  5534.9 1300.42
#Mann=3,-1,0
  4502.8    0.15       0  4974.0    0.05       0  5026.0    0.15       0
Bank Sta=4974,5026
XS Rating Curve= 0
Exp/Cntr=0.3,0.1

Type RM Length L Ch R = 1,109755,419,419,419
BEGIN DESCRIPTION:
Chauga River 220.0
END DESCRIPTION:
XS GIS Cut Line= 3
      1329879.77      1074803.59      1329593.59      1074818.99
      1329042.36      1074939.75
#Sta/Elev= 30
  4713.4 1222.24  4738.5 1219.83  4766.2 1211.23  4782.4 1204.59  4795.4 1195.65
  4800.5 1195.96  4827.0 1182.06  4902.9 1152.68  4913.1 1151.87  4926.1 1147.43
  4936.6 1135.70  4940.9 1133.76  4967.8 1125.02  4974.0 1124.73  4974.5 1123.73
  5026.0 1124.73  5036.5 1124.79  5078.9 1136.56  5105.7 1137.30  5130.6 1148.52
  5157.8 1169.85  5233.7 1217.70  5265.7 1232.00  5303.8 1242.09  5330.0 1244.93
  5354.1 1244.27  5461.6 1232.12  5478.1 1227.55  5522.9 1236.61  5564.3 1235.99
#Mann=3,-1,0
  4713.4    0.15       0  4974.0    0.05       0  5026.0    0.15       0
Bank Sta=4974,5026
XS Rating Curve= 0
Exp/Cntr=0.3,0.1

Type RM Length L Ch R = 1,109336,445,445,445
BEGIN DESCRIPTION:
Chauga River 219.0
END DESCRIPTION:
XS GIS Cut Line= 3
      1329943.05      1074779.49      1329537.52      1074422.16
      1329141.80      1074186.07
#Sta/Elev= 30
  4459.5 1235.55  4560.2 1196.61  4597.1 1177.29  4633.3 1154.07  4664.8 1143.81
  4725.7 1139.54  4826.5 1139.20  4867.2 1136.66  4880.5 1132.65  4962.3 1133.32
  4972.8 1127.32  4973.3 1126.32  5027.2 1127.32  5052.9 1147.02  5085.6 1164.57
  5102.9 1168.41  5124.5 1178.57  5160.2 1175.09  5181.7 1185.40  5189.8 1191.89
  5234.4 1208.29  5255.6 1221.33  5279.3 1228.20  5290.3 1242.97  5299.1 1246.91
  5317.3 1245.49  5333.4 1253.06  5372.8 1263.05  5432.1 1258.26  5460.8 1251.85
#Mann=3,-1,0
  4459.5    0.15       0  4972.8    0.05       0  5027.2    0.15       0
Bank Sta=4972.8,5027.2
XS Rating Curve= 0
Exp/Cntr=0.3,0.1

Type RM Length L Ch R = 1,108891,312,312,312
BEGIN DESCRIPTION:
Chauga River 218.0
END DESCRIPTION:
XS GIS Cut Line= 3
      1329982.21      1074779.46      1329931.58      1074299.22
      1329949.08      1074053.44
#Sta/Elev= 30
  4517.1 1243.79  4561.7 1222.22  4586.8 1207.71  4592.5 1202.95  4603.6 1205.66
  4621.3 1207.54  4639.9 1202.96  4660.3 1193.99  4703.1 1170.05  4749.8 1149.07
  4766.7 1142.67  4784.0 1138.23  4805.3 1136.06  4834.2 1134.16  4861.6 1134.89
  4912.5 1129.86  4932.7 1129.96  4964.6 1125.32  4972.8 1122.05  4973.3 1121.05
  5026.7 1121.05  5027.2 1122.05  5041.9 1128.77  5089.0 1168.55  5106.4 1186.70
  5128.7 1202.32  5151.5 1224.87  5191.0 1247.85  5241.0 1296.86  5246.4 1298.19
#Mann=3,-1,0
  4517.1    0.15       0  4972.8    0.05       0  5027.2    0.15       0
Bank Sta=4972.8,5027.2
XS Rating Curve= 0
Exp/Cntr=0.3,0.1

Type RM Length L Ch R = 1,108579,388,388,388
BEGIN DESCRIPTION:
Chauga River 217.0
END DESCRIPTION:
XS GIS Cut Line= 3
      1330391.90      1074783.08      1330235.99      1074280.61
      1330181.04      1074066.14
#Sta/Elev= 30
  4473.9 1290.40  4584.0 1274.95  4722.9 1232.72  4748.6 1227.36  4768.3 1229.82
  4776.3 1222.11  4782.2 1220.42  4787.9 1208.73  4809.6 1223.94  4848.0 1198.61
  4910.8 1143.70  4917.2 1120.69  4917.9 1124.62  4924.9 1128.31  4934.1 1123.89
  4939.8 1117.02  4941.0 1121.99  4965.5 1119.48  4972.8 1114.57  4973.3 1113.57
  5027.2 1114.57  5034.8 1118.04  5037.9 1123.54  5047.9 1126.06  5091.6 1167.06
  5133.4 1186.46  5153.2 1199.97  5177.2 1228.31  5197.5 1238.40  5221.4 1240.77
#Mann=3,-1,0
  4473.9    0.15       0  4972.8    0.05       0  5027.2    0.15       0
Bank Sta=4972.8,5027.2
XS Rating Curve= 0
Exp/Cntr=0.3,0.1

Type RM Length L Ch R = 1,108191,691,691,691
BEGIN DESCRIPTION:
Chauga River 216.0
END DESCRIPTION:
XS GIS Cut Line= 3
      1330904.04      1074596.33      1330587.93      1074196.11
      1330265.43      1074047.48
#Sta/Elev= 30
  4490.0 1285.57  4512.5 1283.21  4577.5 1289.95  4625.2 1284.86  4684.9 1267.55
  4727.9 1241.79  4755.8 1238.11  4785.4 1217.30  4888.8 1167.84  4927.6 1131.90
  4933.6 1123.27  4939.8 1107.23  4960.8 1097.83  4972.8 1097.83  4973.3 1096.83
  5027.2 1097.83  5038.0 1098.42  5051.1 1108.04  5052.8 1118.71  5060.8 1119.52
  5064.9 1126.84  5138.6 1169.75  5166.3 1173.01  5192.7 1186.05  5213.9 1187.89
  5255.8 1202.41  5268.6 1194.36  5273.5 1207.68  5290.0 1200.64  5355.1 1218.01
#Mann=3,-1,0
  4490.0    0.15       0  4972.8    0.05       0  5027.2    0.15       0
Bank Sta=4972.8,5027.2
XS Rating Curve= 0
Exp/Cntr=0.3,0.1

Type RM Length L Ch R = 1,107500,500,500,500
BEGIN DESCRIPTION:
Chauga River 215.0
END DESCRIPTION:
XS GIS Cut Line= 3
      1331283.61      1074047.46      1331034.02      1073692.04
      1330801.62      1073405.81
#Sta/Elev= 30
  4565.7 1346.36  4688.5 1311.08  4826.5 1198.09  4837.7 1190.35  4845.0 1203.81
  4851.6 1182.74  4876.6 1164.09  4899.5 1160.10  4906.1 1151.22  4920.8 1105.42
  4942.4 1099.32  4943.4 1086.80  4946.6 1079.71  4972.8 1076.74  4973.3 1075.74
  5027.2 1076.74  5034.2 1079.18  5040.0 1089.59  5048.1 1092.87  5048.9 1087.74
  5053.2 1105.11  5056.9 1109.00  5114.6 1151.21  5134.0 1176.06  5170.6 1206.96
  5198.3 1247.90  5248.9 1279.39  5281.1 1286.14  5323.2 1319.52  5368.7 1336.70
#Mann=3,-1,0
  4565.7    0.15       0  4972.8    0.05       0  5027.2    0.15       0
Bank Sta=4972.8,5027.2
XS Rating Curve= 0
Exp/Cntr=0.3,0.1

Type RM Length L Ch R = 1,107000,500,500,500
BEGIN DESCRIPTION:
Chauga River 214.0
END DESCRIPTION:
XS GIS Cut Line= 3
      1331542.69      1073806.49      1331395.60      1073352.84
      1331226.35      1073047.28
#Sta/Elev= 30
  4523.1 1237.01  4546.0 1247.90  4591.4 1246.17  4662.0 1220.38  4663.1 1211.78
  4667.9 1222.83  4712.2 1227.89  4754.8 1221.79  4813.2 1196.81  4837.4 1181.00
  4845.4 1169.72  4860.2 1166.30  4873.0 1132.28  4922.3 1080.71  4950.0 1068.03
  4952.3 1072.40  4972.8 1060.06  4973.3 1059.06  5027.2 1060.06  5055.9 1072.12
  5096.0 1119.82  5108.2 1122.99  5133.0 1170.11  5148.0 1178.44  5158.5 1200.92
  5179.2 1230.49  5204.9 1248.00  5260.5 1302.99  5302.2 1314.78  5349.3 1313.55
#Mann=3,-1,0
  4523.1    0.15       0  4972.8    0.05       0  5027.2    0.15       0
Bank Sta=4972.8,5027.2
XS Rating Curve= 0
Exp/Cntr=0.3,0.1

Type RM Length L Ch R = 1,106500,551,551,551
BEGIN DESCRIPTION:
Chauga River 213.0
END DESCRIPTION:
XS GIS Cut Line= 3
      1331979.48      1073635.31      1331880.69      1073317.93
      1331705.36      1072939.47
#Sta/Elev= 30
  4667.6 1229.12  4681.4 1220.55  4715.4 1211.29  4742.7 1184.54  4776.2 1172.86
  4788.0 1174.08  4820.1 1152.90  4832.5 1151.67  4859.6 1138.92  4866.4 1130.85
  4893.1 1125.90  4916.3 1107.52  4947.8 1063.18  4959.0 1057.16  4966.9 1058.98
  4972.8 1049.04  4973.3 1048.04  5027.2 1049.04  5036.2 1049.29  5054.4 1057.69
  5054.5 1050.68  5057.0 1055.23  5076.9 1056.54  5102.7 1103.69  5134.9 1123.59
  5165.3 1148.02  5217.8 1174.70  5363.8 1204.94  5406.2 1198.67  5417.1 1200.45
#Mann=3,-1,0
  4667.6    0.15       0  4972.8    0.05       0  5027.2    0.15       0
Bank Sta=4972.8,5027.2
XS Rating Curve= 0
Exp/Cntr=0.3,0.1

Type RM Length L Ch R = 1,105949,449,449,449
BEGIN DESCRIPTION:
Chauga River 212.0
END DESCRIPTION:
XS GIS Cut Line= 3
      1332074.98      1073575.03      1332387.05      1073136.54
      1332777.83      1072921.38
#Sta/Elev= 30
  4461.8 1218.30  4516.5 1203.85  4575.2 1175.26  4583.6 1175.41  4632.2 1150.15
  4644.0 1148.40  4654.4 1140.49  4667.9 1140.09  4735.8 1102.46  4747.1 1087.08
  4807.0 1060.20  4848.2 1051.14  4941.0 1043.22  4944.8 1046.37  4972.6 1037.05
  4973.1 1036.05  5027.4 1037.05  5067.5 1041.41  5110.3 1105.41  5120.8 1109.24
  5121.5 1104.52  5123.2 1109.16  5135.6 1110.02  5172.7 1098.39  5179.6 1109.40
  5188.6 1112.60  5202.0 1113.21  5352.1 1164.02  5401.3 1171.13  5446.1 1194.24
#Mann=3,-1,0
  4461.8    0.15       0  4972.6    0.05       0  5027.4    0.15       0
Bank Sta=4972.6,5027.4
XS Rating Curve= 0
Exp/Cntr=0.3,0.1

Type RM Length L Ch R = 1,105500,389,389,389
BEGIN DESCRIPTION:
Chauga River 211.0
END DESCRIPTION:
XS GIS Cut Line= 3
      1332066.84      1073654.03      1332457.85      1073559.83
      1332663.31      1073521.48
#Sta/Elev= 30
  4597.8 1237.08  4636.6 1226.60  4651.3 1216.92  4698.8 1197.73  4776.6 1152.78
  4864.0 1090.02  4896.4 1074.82  4913.7 1051.67  4922.8 1055.04  4936.9 1051.91
  4939.7 1035.41  4942.1 1035.62  4946.2 1047.15  4948.8 1045.58  4956.4 1031.99
  4972.6 1030.56  4973.1 1029.56  5027.4 1030.56  5031.7 1041.02  5036.7 1042.78
  5040.7 1039.56  5084.4 1072.21  5098.1 1093.55  5119.2 1111.58  5130.5 1116.87
  5147.6 1132.49  5152.4 1133.70  5158.1 1140.23  5176.5 1153.45  5209.0 1158.80
#Mann=3,-1,0
  4597.8    0.15       0  4972.6    0.05       0  5027.4    0.15       0
Bank Sta=4972.6,5027.4
XS Rating Curve= 0
Exp/Cntr=0.3,0.1

Type RM Length L Ch R = 1,105111,611,611,611
BEGIN DESCRIPTION:
Chauga River 210.0
END DESCRIPTION:
XS GIS Cut Line= 3
      1332506.67      1074211.37      1332670.01      1073807.55
      1332711.53      1073500.35
#Sta/Elev= 30
  4564.4 1209.45  4595.1 1205.35  4609.0 1209.10  4637.0 1204.69  4668.3 1209.48
  4710.5 1203.12  4759.2 1182.13  4772.3 1174.12  4786.1 1154.37  4808.7 1145.00
  4814.4 1146.44  4834.8 1126.39  4843.0 1124.05  4868.3 1106.10  4902.6 1061.81
  4903.5 1065.31  4919.2 1056.02  4939.7 1034.80  4972.4 1024.14  4972.9 1023.14
  5027.6 1024.14  5043.7 1032.39  5052.1 1030.00  5072.7 1044.21  5098.5 1051.59
  5107.1 1058.00  5128.1 1090.13  5139.4 1090.65  5151.6 1100.19  5310.0 1167.33
#Mann=3,-1,0
  4564.4    0.15       0  4972.4    0.05       0  5027.6    0.15       0
Bank Sta=4972.4,5027.6
XS Rating Curve= 0
Exp/Cntr=0.3,0.1

Type RM Length L Ch R = 1,104500,500,500,500
BEGIN DESCRIPTION:
Chauga River 209.0
END DESCRIPTION:
XS GIS Cut Line= 3
      1333323.07      1073801.65      1333198.54      1073511.55
      1332991.67      1073256.37
#Sta/Elev= 30
  4684.3 1138.70  4747.1 1108.68  4773.0 1100.80  4790.9 1085.42  4804.9 1085.30
  4834.0 1066.73  4876.6 1047.11  4887.6 1028.48  4898.4 1019.84  4900.2 1022.92
  4909.0 1011.86  4940.4 1012.87  4956.6 1023.97  4972.4 1011.86  4972.9 1010.86
  5027.6 1011.86  5028.0 1020.09  5041.2 1022.00  5041.5 1018.58  5044.4 1024.76
  5051.7 1025.45  5080.6 1048.38  5097.2 1073.54  5125.4 1080.37  5173.7 1112.79
  5188.3 1135.14  5220.9 1145.22  5232.9 1160.82  5258.9 1165.71  5328.5 1201.63
#Mann=3,-1,0
  4684.3    0.15       0  4972.4    0.05       0  5027.6    0.15       0
Bank Sta=4972.4,5027.6
XS Rating Curve= 0
Exp/Cntr=0.3,0.1

Type RM Length L Ch R = 1,104000,500,500,500
BEGIN DESCRIPTION:
Chauga River 208.0
END DESCRIPTION:
XS GIS Cut Line= 3
      1333359.24      1073810.65      1333657.89      1073567.53
      1333868.30      1073181.10
#Sta/Elev= 30
  4614.9 1138.85  4731.3 1120.70  4758.2 1107.03  4809.5 1090.32  4823.2 1079.04
  4841.9 1074.32  4865.0 1060.88  4882.7 1043.36  4924.2 1025.73  4950.4 1019.89
  4952.6 1012.14  4972.4 1001.85  4972.9 1000.85  5027.6 1001.85  5034.6 1006.37
  5046.5 1003.99  5058.1 1027.36  5062.0 1015.19  5062.3 1009.99  5065.3 1018.42
  5085.3 1042.57  5144.3 1087.30  5198.6 1137.88  5248.0 1165.59  5296.8 1178.79
  5310.4 1177.10  5355.1 1200.72  5378.2 1207.26  5402.0 1206.18  5440.0 1189.02
#Mann=3,-1,0
  4614.9    0.15       0  4972.4    0.05       0  5027.6    0.15       0
Bank Sta=4972.4,5027.6
XS Rating Curve= 0
Exp/Cntr=0.3,0.1

Type RM Length L Ch R = 1,103500,500,500,500
BEGIN DESCRIPTION:
Chauga River 207.0
END DESCRIPTION:
XS GIS Cut Line= 3
      1334112.33      1074048.64      1334148.73      1073648.59
      1334175.60      1073232.26
#Sta/Elev= 30
  4598.3 1147.85  4663.0 1110.56  4704.4 1091.48  4765.4 1067.27  4779.0 1067.34
  4795.6 1056.63  4907.9 1021.44  4923.1 1011.45  4951.7 1001.53  4967.1 1006.72
  4969.7 1004.21  4972.4  995.38  4972.9  994.38  5027.6  995.38  5053.0 1013.28
  5056.1  998.56  5056.6 1009.67  5062.2 1026.78  5071.9 1007.85  5072.8 1009.44
  5072.9 1004.01  5073.5 1021.43  5077.6 1036.21  5096.9 1057.49  5126.9 1077.19
  5160.1 1106.90  5181.1 1116.63  5294.8 1155.21  5343.5 1166.45  5417.2 1171.04
#Mann=3,-1,0
  4598.3    0.15       0  4972.4    0.05       0  5027.6    0.15       0
Bank Sta=4972.4,5027.6
XS Rating Curve= 0
Exp/Cntr=0.3,0.1

Type RM Length L Ch R = 1,103000,500,500,500
BEGIN DESCRIPTION:
Chauga River 206.0
END DESCRIPTION:
XS GIS Cut Line= 3
      1334627.46      1073970.38      1334647.40      1073678.25
      1334684.70      1073229.30
#Sta/Elev= 30
  4707.2 1144.42  4734.3 1125.83  4736.2 1139.94  4742.3 1122.96  4756.9 1114.78
  4815.4 1101.41  4913.5 1054.23  4971.9 1001.69  4972.4  988.84  4972.9  987.84
  5027.6  988.84  5039.0  998.45  5052.2 1000.63  5054.9  999.23  5056.0  991.80
  5070.5 1018.22  5070.7  997.66  5073.5 1015.80  5078.7 1023.02  5104.2 1042.42
  5111.7 1057.18  5122.9 1067.42  5149.9 1082.75  5211.4 1093.50  5289.4 1085.38
  5355.9 1118.63  5378.2 1141.03  5406.6 1141.30  5422.6 1153.64  5450.5 1161.82
#Mann=3,-1,0
  4707.2    0.15       0  4972.4    0.05       0  5027.6    0.15       0
Bank Sta=4972.4,5027.6
XS Rating Curve= 0
Exp/Cntr=0.3,0.1

Type RM Length L Ch R = 1,102500,570,570,570
BEGIN DESCRIPTION:
Chauga River 205.0
END DESCRIPTION:
XS GIS Cut Line= 3
      1334696.75      1073997.45      1335094.26      1073808.12
      1335422.72      1073702.24
#Sta/Elev= 30
  4559.7 1158.52  4602.4 1142.66  4629.6 1128.61  4658.6 1109.17  4685.1 1096.43
  4721.6 1087.95  4786.6 1079.66  4842.3 1056.81  4850.8 1056.14  4857.1 1048.53
  4897.9 1031.42  4914.4 1018.98  4935.1  996.33  4961.3  980.89  4972.4  978.61
  4972.9  977.61  5027.6  978.61  5034.3  984.19  5052.0  988.80  5052.4  991.99
  5073.2 1031.45  5074.1 1035.84  5082.4 1043.17  5106.0 1079.66  5140.1 1100.40
  5155.8 1105.39  5191.9 1127.80  5271.7 1158.88  5311.5 1168.60  5345.1 1169.67
#Mann=3,-1,0
  4559.7    0.15       0  4972.4    0.05       0  5027.6    0.15       0
Bank Sta=4972.4,5027.6
XS Rating Curve= 0
Exp/Cntr=0.3,0.1

Type RM Length L Ch R = 1,101930,519,519,519
BEGIN DESCRIPTION:
Chauga River 204.0
END DESCRIPTION:
XS GIS Cut Line= 3
      1334913.67      1074836.71      1335280.15      1074337.49
      1335455.87      1074158.95
#Sta/Elev= 30
  4380.7 1245.67  4394.6 1236.83  4414.9 1238.61  4450.1 1222.25  4487.9 1217.04
  4499.1 1208.01  4560.2 1188.90  4632.0 1148.18  4662.6 1141.06  4671.9 1133.80
  4682.5 1137.29  4687.1 1129.71  4847.9 1037.93  4865.7 1023.40  4912.3  998.41
  4923.4  987.02  4937.8  988.76  4962.6  971.71  4972.4  971.49  4972.9  970.49
  5027.6  971.49  5043.1  971.49  5072.6 1016.34  5081.0 1002.93  5081.7  975.57
  5084.2 1005.28  5100.5 1024.15  5115.2 1051.70  5189.9 1087.37  5250.5 1096.66
#Mann=3,-1,0
  4380.7    0.15       0  4972.4    0.05       0  5027.6    0.15       0
Bank Sta=4972.4,5027.6
XS Rating Curve= 0
Exp/Cntr=0.3,0.1

Type RM Length L Ch R = 1,101411,411,411,411
BEGIN DESCRIPTION:
Chauga River 203.0
END DESCRIPTION:
XS GIS Cut Line= 3
      1336136.75      1074731.32      1335728.09      1074354.47
      1335495.03      1074068.51
#Sta/Elev= 30
  4444.1 1174.41  4476.1 1176.50  4575.2 1164.21  4590.0 1165.95  4728.4 1139.21
  4775.3 1139.90  4805.7 1124.67  4835.6 1119.60  4880.6 1093.51  4900.3 1077.72
  4928.7 1038.38  4941.5  967.06  4946.2  995.81  4952.7  973.35  4960.3  977.20
  4964.5  963.58  4972.2  962.50  4972.7  961.50  5027.8  962.50  5036.3  970.11
  5067.1  976.32  5067.9  965.02  5092.8  978.79  5129.5  984.04  5216.1 1017.56
  5282.1 1072.73  5309.1 1084.87  5320.2 1083.21  5337.6 1104.57  5368.9 1114.68
#Mann=3,-1,0
  4444.1    0.15       0  4972.2    0.05       0  5027.8    0.15       0
Bank Sta=4972.2,5027.8
XS Rating Curve= 0
Exp/Cntr=0.3,0.1

Type RM Length L Ch R = 1,101000,500,500,500
BEGIN DESCRIPTION:
Chauga River 202.0
END DESCRIPTION:
XS GIS Cut Line= 3
      1336377.74      1074260.75      1335925.77      1073999.98
      1335576.39      1073811.88
#Sta/Elev= 30
  4478.2 1117.56  4541.7 1095.34  4638.6 1034.67  4707.9 1004.31  4717.6  983.51
  4723.7 1012.21  4780.5 1017.07  4809.0 1009.02  4838.2 1015.40  4880.6 1004.79
  4905.8 1005.03  4925.1  971.77  4925.3  963.41  4926.6  987.01  4950.5  964.25
  4972.2  956.32  4972.7  955.32  5027.8  956.32  5040.8  968.06  5072.9  958.11
  5080.4  977.19  5096.2  975.21  5099.1  956.79  5103.9  986.17  5109.0  998.27
  5136.7 1016.59  5173.5 1062.24  5216.7 1072.89  5308.3 1135.49  5396.8 1168.32
#Mann=3,-1,0
  4478.2    0.15       0  4972.2    0.05       0  5027.8    0.15       0
Bank Sta=4972.2,5027.8
XS Rating Curve= 0
Exp/Cntr=0.3,0.1

Type RM Length L Ch R = 1,100500,536,536,536
BEGIN DESCRIPTION:
Chauga River 201.0
END DESCRIPTION:
XS GIS Cut Line= 3
      1336630.76      1074209.52      1336356.80      1073774.15
      1336224.08      1073540.75
#Sta/Elev= 30
  4485.6 1150.74  4541.0 1135.33  4561.6 1124.02  4580.9 1117.22  4634.6 1105.64
  4686.1 1085.98  4701.3 1082.47  4714.6 1075.80  4726.4 1073.23  4864.2 1005.72
  4897.4  984.74  4912.2  970.48  4928.5  958.46  4947.0  956.19  4963.0  949.70
  4971.8  949.70  4972.3  948.70  5028.2  949.70  5031.7  954.51  5039.4  950.12
  5053.1  955.08  5058.2  955.00  5059.7  959.16  5064.2  955.29  5078.0  954.68
  5129.8  965.12  5216.2  997.82  5256.9 1009.57  5265.8  983.34  5268.5  982.13
#Mann=3,-1,0
  4485.6    0.15       0  4971.8    0.05       0  5028.2    0.15       0
Bank Sta=4971.8,5028.2
XS Rating Curve= 0
Exp/Cntr=0.3,0.1

Type RM Length L Ch R = 1,99964,464,464,464
BEGIN DESCRIPTION:
Chauga River 200.0
END DESCRIPTION:
XS GIS Cut Line= 3
      1337188.09      1073623.31      1336777.04      1073465.23
      1336215.07      1073511.84
#Sta/Elev= 30
  4559.6 1240.46  4569.7 1223.94  4615.3 1199.07  4627.2 1182.39  4660.1 1149.46
  4705.1 1121.39  4761.1 1100.41  4777.5 1087.90  4825.3 1063.84  4845.2 1061.81
  4855.6 1067.83  4866.5 1059.46  4886.0 1055.17  4898.9 1046.90  4924.9 1020.15
  4947.9  981.09  4960.7  972.07  4966.2  951.37  4971.8  943.84  4972.3  942.84
  5028.2  943.84  5036.7  948.64  5043.6  946.01  5078.7  951.79  5252.4  956.69
  5381.0  966.34  5449.3  988.12  5526.9 1005.22  5556.8 1006.79  5563.9 1001.71
#Mann=3,-1,0
  4559.6    0.15       0  4971.8    0.05       0  5028.2    0.15       0
Bank Sta=4971.8,5028.2
XS Rating Curve= 0
Exp/Cntr=0.3,0.1

Type RM Length L Ch R = 1,99500,500,500,500
BEGIN DESCRIPTION:
Chauga River 199.0
END DESCRIPTION:
XS GIS Cut Line= 3
      1337371.82      1073328.07      1336939.28      1073039.80
      1336443.98      1072689.42
#Sta/Elev= 30
  4480.2 1224.31  4520.4 1203.87  4528.2 1191.28  4531.4 1198.50  4558.5 1185.31
  4603.5 1177.54  4655.2 1149.58  4701.1 1135.30  4725.2 1105.17  4763.5 1081.14
  4765.8 1074.58  4830.3 1033.45  4844.1 1018.56  4859.0 1013.74  4869.5 1000.89
  4899.4  991.25  4902.6  976.20  4907.6  967.84  4922.1  956.02  4971.8  940.58
  4972.3  939.58  5028.2  940.58  5073.7  949.24  5179.2  954.20  5237.5  970.45
  5330.8 1029.66  5375.5 1040.82  5415.7 1063.97  5532.3 1153.19  5606.7 1201.29
#Mann=3,-1,0
  4480.2    0.15       0  4971.8    0.05       0  5028.2    0.15       0
Bank Sta=4971.8,5028.2
XS Rating Curve= 0
Exp/Cntr=0.3,0.1

Type RM Length L Ch R = 1,99000,500,500,500
BEGIN DESCRIPTION:
Chauga River 198.0
END DESCRIPTION:
XS GIS Cut Line= 3
      1337435.12      1072830.43      1337103.35      1072576.32
      1336627.72      1072236.93
#Sta/Elev= 30
  4582.1 1107.61  4618.4 1091.48  4658.8 1064.55  4663.7 1057.43  4698.7 1028.84
  4733.2  992.30  4768.9  972.93  4782.9  967.50  4784.8  969.01  4787.9  980.76
  4792.0  971.82  4792.8  964.69  4872.0  944.07  4917.8  947.61  4971.8  936.71
  4972.3  935.71  5028.2  936.71  5028.6  957.10  5029.4  957.92  5042.9  937.25
  5073.8  972.97  5250.7 1063.44  5254.7 1068.94  5254.8 1074.48  5277.1 1077.74
  5324.0 1099.11  5403.0 1149.17  5436.7 1159.18  5536.1 1175.83  5584.3 1199.41
#Mann=3,-1,0
  4582.1    0.15       0  4971.8    0.05       0  5028.2    0.15       0
Bank Sta=4971.8,5028.2
XS Rating Curve= 0
Exp/Cntr=0.3,0.1

Type RM Length L Ch R = 1,98500,500,500,500
BEGIN DESCRIPTION:
Chauga River 197.0
END DESCRIPTION:
XS GIS Cut Line= 3
      1337540.53      1072682.77      1337479.99      1072267.15
      1337417.03      1071932.73
#Sta/Elev= 30
  4580.0 1058.32  4615.9 1039.75  4618.1 1029.60  4625.6 1051.75  4705.4 1023.16
  4818.4  958.67  4843.8  951.58  4912.8  944.25  4934.2  946.63  4952.6  935.43
  4971.8  935.43  4972.3  934.43  5028.2  935.43  5031.7  943.20  5043.6  935.60
  5056.4  953.72  5058.2  943.39  5060.9  936.71  5078.2  967.24  5094.8  986.21
  5120.7  994.66  5123.3 1001.93  5162.2 1029.06  5175.2 1044.88  5200.8 1057.34
  5218.9 1071.22  5232.9 1095.17  5259.8 1104.13  5294.0 1139.32  5340.3 1164.15
#Mann=3,-1,0
  4580.0    0.15       0  4971.8    0.05       0  5028.2    0.15       0
Bank Sta=4971.8,5028.2
XS Rating Curve= 0
Exp/Cntr=0.3,0.1

Type RM Length L Ch R = 1,98000,500,500,500
BEGIN DESCRIPTION:
Chauga River 196.0
END DESCRIPTION:
XS GIS Cut Line= 3
      1338206.30      1072288.78      1337876.49      1071995.27
      1337459.24      1071854.99
#Sta/Elev= 30
  4558.5 1141.24  4571.6 1146.81  4631.3 1120.69  4641.7 1122.96  4672.7 1104.75
  4710.2 1095.72  4724.0 1075.93  4736.6 1077.48  4799.6 1035.79  4822.8 1032.72
  4839.5 1022.15  4871.9  995.99  4907.7  956.23  4923.2  944.97  4971.8  930.25
  4972.3  929.25  5028.2  930.25  5035.7  940.90  5040.4  931.38  5048.4  937.13
  5063.7  958.09  5088.4  976.63  5116.5 1009.76  5146.0 1015.96  5213.1 1044.82
  5281.1 1057.52  5310.5 1069.82  5356.1 1100.44  5392.6 1110.24  5440.2 1136.72
#Mann=3,-1,0
  4558.5    0.15       0  4971.8    0.05       0  5028.2    0.15       0
Bank Sta=4971.8,5028.2
XS Rating Curve= 0
Exp/Cntr=0.3,0.1

Type RM Length L Ch R = 1,97500,620,620,620
BEGIN DESCRIPTION:
Chauga River 195.0
END DESCRIPTION:
XS GIS Cut Line= 3
      1338353.92      1071943.57      1338160.00      1071599.56
      1337926.12      1071208.46
#Sta/Elev= 30
  4605.1 1138.32  4626.4 1133.11  4661.0 1112.53  4675.3 1098.53  4724.2 1076.71
  4748.7 1060.15  4805.5 1041.75  4821.1 1022.99  4839.1 1006.52  4846.7 1005.27
  4878.3  974.15  4917.5  949.06  4932.8  951.62  4949.0  931.30  4957.6  932.78
  4971.8  925.15  4972.3  924.15  5028.2  925.15  5051.7  931.34  5063.8  951.57
  5084.8  963.63  5107.9  985.08  5119.7 1005.84  5154.4 1012.95  5207.5 1040.11
  5256.2 1082.27  5319.0 1106.50  5360.6 1110.62  5395.3 1134.70  5455.7 1157.82
#Mann=3,-1,0
  4605.1    0.15       0  4971.8    0.05       0  5028.2    0.15       0
Bank Sta=4971.8,5028.2
XS Rating Curve= 0
Exp/Cntr=0.3,0.1

Type RM Length L Ch R = 1,96880,455,455,455
BEGIN DESCRIPTION:
Chauga River 194.0
END DESCRIPTION:
XS GIS Cut Line= 3
      1338522.60      1071762.82      1338651.85      1071244.59
      1338748.53      1070910.29
#Sta/Elev= 30
  4465.9 1108.00  4618.4 1061.09  4624.4 1064.22  4636.1 1055.35  4692.6 1042.39
  4882.2  978.37  4892.0  969.16  4907.2  965.87  4936.4  939.32  4937.2  930.57
  4950.7  923.27  4971.8  920.51  4972.3  919.51  5028.2  920.51  5043.3  925.73
  5044.5  920.51  5051.6  927.72  5075.7  928.26  5087.9  945.18  5120.5  962.19
  5154.5  989.85  5163.5 1001.97  5189.9 1017.92  5223.3 1045.87  5246.9 1080.04
  5258.4 1081.85  5269.5 1099.49  5290.5 1107.81  5295.9 1114.81  5348.0 1122.48
#Mann=3,-1,0
  4465.9    0.15       0  4971.8    0.05       0  5028.2    0.15       0
Bank Sta=4971.8,5028.2
XS Rating Curve= 0
Exp/Cntr=0.3,0.1

Type RM Length L Ch R = 1,96425,335,335,335
BEGIN DESCRIPTION:
Chauga River 193.0
END DESCRIPTION:
XS GIS Cut Line= 3
      1338561.77      1071937.52      1338847.86      1071624.18
      1339010.65      1071452.49
#Sta/Elev= 30
  4575.7 1123.98  4618.0 1111.67  4668.1 1091.16  4705.4 1067.61  4725.4 1059.21
  4739.0 1050.32  4745.6 1038.01  4750.7 1043.37  4767.2 1035.05  4794.6 1029.12
  4802.2 1019.13  4809.7 1012.70  4818.2 1011.49  4849.7  990.84  4866.5  982.48
  4887.1  958.15  4926.8  942.30  4956.3  918.67  4971.8  916.75  4972.3  915.75
  5028.2  916.75  5029.0  921.77  5033.3  919.94  5042.7  924.49  5045.1  933.95
  5055.1  925.95  5070.3  955.63  5094.3  974.93  5156.9 1005.58  5236.6 1024.07
#Mann=3,-1,0
  4575.7    0.15       0  4971.8    0.05       0  5028.2    0.15       0
Bank Sta=4971.8,5028.2
XS Rating Curve= 0
Exp/Cntr=0.3,0.1

Type RM Length L Ch R = 1,96090,693,693,693
BEGIN DESCRIPTION:
Chauga River 192.0
END DESCRIPTION:
XS GIS Cut Line= 3
      1339272.71      1072136.31      1339159.41      1071670.59
      1339055.81      1071362.12
#Sta/Elev= 30
  4520.7 1099.42  4566.5 1085.27  4637.1 1069.33  4654.9 1057.61  4675.0 1050.15
  4696.1 1047.54  4737.8 1031.83  4797.9  998.28  4805.9  996.37  4811.5  988.26
  4827.3  979.33  4857.8  970.51  4867.5  961.01  4900.9  953.32  4915.7  945.49
  4930.5  937.07  4943.5  919.58  4949.4  915.40  4971.8  911.68  4972.3  910.68
  5028.2  911.68  5037.5  917.60  5092.6  926.20  5113.9  939.07  5122.9  947.83
  5180.2  979.68  5208.8 1009.86  5233.4 1014.14  5275.0 1040.73  5325.4 1058.98
#Mann=3,-1,0
  4520.7    0.15       0  4971.8    0.05       0  5028.2    0.15       0
Bank Sta=4971.8,5028.2
XS Rating Curve= 0
Exp/Cntr=0.3,0.1

Type RM Length L Ch R = 1,95397,567,567,567
BEGIN DESCRIPTION:
Chauga River 191.0
END DESCRIPTION:
XS GIS Cut Line= 3
      1339971.63      1071621.23      1339691.81      1071232.58
      1339384.23      1070928.38
#Sta/Elev= 30
  4521.1 1027.48  4577.0 1021.59  4581.2 1007.65  4582.5 1020.80  4704.3  978.46
  4787.8  961.04  4872.2  928.72  4916.8  917.70  4949.4  914.13  4971.8  905.21
  4972.3  904.21  5028.2  905.21  5040.3  909.95  5063.0  910.48  5064.5  905.36
  5064.6  908.33  5072.3  912.29  5074.2  917.35  5076.6  910.53  5076.9  918.31
  5082.4  915.49  5114.2  942.91  5152.8  968.39  5175.3  988.77  5184.0  992.45
  5201.6  994.20  5245.7 1007.67  5310.1 1006.47  5375.8 1025.57  5432.6 1034.31
#Mann=3,-1,0
  4521.1    0.15       0  4971.8    0.05       0  5028.2    0.15       0
Bank Sta=4971.8,5028.2
XS Rating Curve= 0
Exp/Cntr=0.3,0.1

Type RM Length L Ch R = 1,94830,452,452,452
BEGIN DESCRIPTION:
Chauga River 190.0
END DESCRIPTION:
XS GIS Cut Line= 3
      1340471.68      1070945.81      1340098.30      1070841.40
      1339754.72      1070734.93
#Sta/Elev= 30
  4612.3  985.64  4675.2 1000.69  4727.8  995.25  4760.5  984.81  4813.8  961.46
  4822.6  956.45  4826.7  945.62  4828.0  946.79  4829.3  952.61  4912.3  914.92
  4913.1  916.81  4915.2  912.32  4936.2  908.62  4949.6  909.06  4960.6  905.00
  4963.2  898.21  4969.7  897.94  4970.2  896.94  5030.3  897.94  5039.5  901.91
  5045.2  897.94  5057.1  907.44  5062.4  908.28  5068.4  906.02  5109.1  907.27
  5182.9  921.55  5213.6  933.55  5297.5  974.06  5335.6  988.56  5359.7  994.38
#Mann=3,-1,0
  4612.3    0.15       0  4969.7    0.05       0  5030.3    0.15       0
Bank Sta=4969.7,5030.3
XS Rating Curve= 0
Exp/Cntr=0.3,0.1

Type RM Length L Ch R = 1,94378,378,378,378
BEGIN DESCRIPTION:
Chauga River 189.0
END DESCRIPTION:
XS GIS Cut Line= 3
      1340426.47      1070367.41      1340168.26      1070408.79
      1339769.74      1070575.29
#Sta/Elev= 30
  4738.5 1004.77  4780.2 1001.75  4781.0 1006.67  4782.0 1001.68  4821.0  987.99
  4863.4  965.04  4875.5  964.51  4878.2  968.47  4878.8  960.75  4879.6  960.03
  4889.8  958.17  4928.0  931.76  4932.8  924.10  4937.2  904.65  4939.1  904.56
  4948.2  920.74  4958.4  904.58  4960.9  897.78  4969.7  896.28  4970.2  895.28
  5030.3  896.28  5044.3  913.06  5044.7  910.07  5052.1  902.64  5089.3  902.50
  5202.2  927.79  5221.3  927.21  5342.2  959.22  5372.0  964.15  5431.9  967.60
#Mann=3,-1,0
  4738.5    0.15       0  4969.7    0.05       0  5030.3    0.15       0
Bank Sta=4969.7,5030.3
XS Rating Curve= 0
Exp/Cntr=0.3,0.1

Type RM Length L Ch R = 1,94000,500,500,500
BEGIN DESCRIPTION:
Chauga River 188.0
END DESCRIPTION:
XS GIS Cut Line= 3
      1340518.68      1070059.53      1340137.62      1070034.21
      1339570.99      1069966.15
#Sta/Elev= 30
  4618.1  958.13  4619.8  958.68  4622.6  980.41  4623.1  967.39  4625.3  960.95
  4659.8  971.57  4687.8  970.38  4809.2  926.41  4835.8  920.93  4838.5  927.25
  4840.0  919.95  4861.1  915.55  4865.1  908.15  4866.0  914.90  4921.3  908.98
  4937.7  904.60  4938.4  898.20  4941.1  903.99  4969.7  896.28  4970.2  895.28
  5030.3  896.28  5058.7  907.53  5198.8  902.84  5200.5  915.73  5205.6  925.59
  5208.9  904.26  5289.8  905.07  5424.3  964.59  5491.5  983.13  5570.7  992.88
#Mann=3,-1,0
  4618.1    0.15       0  4969.7    0.05       0  5030.3    0.15       0
Bank Sta=4969.7,5030.3
XS Rating Curve= 0
Exp/Cntr=0.3,0.1

Type RM Length L Ch R = 1,93500,500,500,500
BEGIN DESCRIPTION:
Chauga River 187.0
END DESCRIPTION:
XS GIS Cut Line= 3
      1340663.28      1069696.83      1340351.21      1069596.50
      1339777.64      1069428.73
#Sta/Elev= 30
  4672.2  956.12  4744.8  940.10  4791.2  936.86  4792.7  937.28  4792.9  945.26
  4795.2  936.95  4876.2  917.89  4883.1  910.27  4906.0  911.79  4924.2  902.94
  4928.5  907.56  4933.3  900.26  4969.5  890.29  4970.0  889.29  5030.5  890.29
  5055.3  896.53  5073.2  890.29  5075.1  900.58  5241.5  923.92  5324.3  948.29
  5337.6  959.28  5359.5  958.72  5367.4  975.03  5370.1  996.41  5375.7  962.32
  5485.1  965.11  5491.2  996.41  5499.3  962.50  5547.6  950.91  5597.6  973.62
#Mann=3,-1,0
  4672.2    0.15       0  4969.5    0.05       0  5030.5    0.15       0
Bank Sta=4969.5,5030.5
XS Rating Curve= 0
Exp/Cntr=0.3,0.1

Type RM Length L Ch R = 1,93000,500,500,500
BEGIN DESCRIPTION:
Chauga River 186.0
END DESCRIPTION:
XS GIS Cut Line= 3
      1340720.51      1069648.61      1340623.04      1069214.52
      1340569.90      1068862.41
#Sta/Elev= 30
  4555.1  974.90  4616.8  962.67  4713.4  929.54  4787.8  916.16  4798.9  909.63
  4807.1  913.74  4950.6  899.75  4969.5  890.07  4970.0  889.07  5030.5  890.07
  5065.6  902.92  5098.8  931.90  5107.4  890.47  5113.0  933.34  5115.2  932.68
  5118.3  897.95  5119.2  899.32  5121.1  917.99  5122.0  903.62  5123.8  917.22
  5128.4  932.18  5130.3  963.87  5179.0  996.20  5242.9 1018.65  5252.3 1029.94
  5256.2 1045.54  5257.8 1029.97  5262.5 1028.03  5262.8 1022.71  5356.1 1038.17
#Mann=3,-1,0
  4555.1    0.15       0  4969.5    0.05       0  5030.5    0.15       0
Bank Sta=4969.5,5030.5
XS Rating Curve= 0
Exp/Cntr=0.3,0.1
