HEC-RAS study Chauga River.prj: Chauga River Limited Detail Study

--- Chauga River.g01 (geometry) --- (continued)

Type RM Length L Ch R = 1,92500,656,656,656
BEGIN DESCRIPTION:
Chauga River 185.0
END DESCRIPTION:
XS GIS Cut Line= 3
      1341142.26      1069705.82      1341122.85      1069222.71
      1341106.11      1068951.53
#Sta/Elev= 30
  4516.5  988.51  4568.4  989.54  4652.1  964.20  4706.1  953.39  4782.2  943.59
  4873.3  912.59  4879.7  911.04  4882.6  913.80  4887.6  909.74  4936.1  896.29
  4968.7  892.09  4969.5  888.07  4970.0  887.07  5030.5  888.07  5059.0  894.93
  5060.0  893.62  5060.6  889.04  5060.8  893.71  5076.7  901.59  5078.6  896.82
  5101.5  925.17  5113.3  933.60  5196.0  971.43  5217.7  978.69  5218.5  989.23
  5230.1  984.18  5232.2  992.40  5233.9  985.24  5235.9  985.02  5271.7  995.88
#Mann=3,-1,0
  4516.5    0.15       0  4969.5    0.05       0  5030.5    0.15       0
Bank Sta=4969.5,5030.5
XS Rating Curve= 0
Exp/Cntr=0.3,0.1

Type RM Length L Ch R = 1,91844,423,423,423
BEGIN DESCRIPTION:
Chauga River 184.0
END DESCRIPTION:
XS GIS Cut Line= 3
      1342223.76      1069662.50      1341680.90      1069007.39
      1341464.61      1068797.92
#Sta/Elev= 30
  4149.2  995.61  4228.9  992.90  4281.9  982.80  4352.8  958.26  4447.8  907.41
  4475.0  902.95  4527.6  902.16  4536.6  911.64  4538.1  904.20  4541.7  901.76
  4783.5  906.80  4879.0  904.09  4924.3  895.30  4925.3  897.86  4925.6  909.84
  4932.6  898.43  4969.5  887.54  4970.0  886.54  5030.5  887.54  5051.8  887.54
  5065.4  904.36  5074.9  894.14  5090.3  896.02  5212.3  929.54  5229.6  938.77
  5254.0  944.71  5258.6  939.99  5266.9  960.08  5267.8  941.74  5301.1  947.05
#Mann=3,-1,0
  4149.2    0.15       0  4969.5    0.05       0  5030.5    0.15       0
Bank Sta=4969.5,5030.5
XS Rating Curve= 0
Exp/Cntr=0.3,0.1

Type RM Length L Ch R = 1,91421,363,363,363
BEGIN DESCRIPTION:
Chauga River 183.0
END DESCRIPTION:
XS GIS Cut Line= 3
      1342627.43      1068665.35      1342014.04      1068779.94
      1341425.45      1068776.82
#Sta/Elev= 30
  4376.0  987.75  4381.3  990.84  4382.7  984.98  4387.0  980.96  4577.2  925.88
  4671.6  925.28  4673.0  912.46  4673.1  917.95  4681.2  923.96  4759.1  923.58
  4888.0  902.32  4896.8  910.11  4897.5  916.83  4904.1  901.12  4945.6  883.31
  4969.5  883.13  4970.0  882.13  5030.5  883.13  5075.3  894.63  5083.3  906.65
  5105.1  892.84  5309.9  902.71  5341.5  924.62  5352.4  903.12  5392.5  908.73
  5394.7  903.93  5403.3  911.17  5444.5  926.05  5506.4  943.93  5588.6  956.25
#Mann=3,-1,0
  4376.0    0.15       0  4969.5    0.05       0  5030.5    0.15       0
Bank Sta=4969.5,5030.5
XS Rating Curve= 0
Exp/Cntr=0.3,0.1

Type RM Length L Ch R = 1,91058,558,558,558
BEGIN DESCRIPTION:
Chauga River 182.0
END DESCRIPTION:
XS GIS Cut Line= 3
      1342094.25      1068468.33      1341741.17      1068563.94
      1341395.32      1068685.24
#Sta/Elev= 30
  4634.2  945.68  4659.7  943.81  4725.3  946.63  4749.0  944.92  4754.6  940.26
  4761.6  943.28  4789.3  938.82  4874.7  921.76  4930.0  895.11  4930.5  898.32
  4937.9  892.50  4955.2  893.63  4966.5  883.41  4969.5  882.98  4970.0  881.98
  5030.5  882.98  5039.6  885.89  5042.6  902.19  5045.1  910.51  5048.8  888.86
  5060.2  888.33  5104.2  895.23  5115.2  923.90  5127.0  903.52  5133.6  894.78
  5143.8  894.50  5212.2  925.47  5272.4  949.32  5324.8  965.03  5366.5  970.97
#Mann=3,-1,0
  4634.2    0.15       0  4969.5    0.05       0  5030.5    0.15       0
Bank Sta=4969.5,5030.5
XS Rating Curve= 0
Exp/Cntr=0.3,0.1

Type RM Length L Ch R = 1,90500,500,500,500
BEGIN DESCRIPTION:
Chauga River 181.0
END DESCRIPTION:
XS GIS Cut Line= 3
      1342187.61      1068180.95      1341858.25      1068054.23
      1341536.94      1067949.00
#Sta/Elev= 30
  4647.1  960.44  4704.0  943.33  4774.2  929.26  4847.6  906.47  4852.5  915.63
  4856.2  905.62  4879.1  899.75  4944.7  895.11  4969.5  880.42  4970.0  879.42
  5030.5  880.42  5040.6  888.82  5041.4  882.11  5042.2  881.85  5056.5  890.06
  5062.5  914.37  5074.8  906.69  5104.3  926.45  5131.9  939.35  5155.8  943.66
  5156.5  944.09  5156.6  948.44  5174.2  947.11  5203.5  973.37  5204.9  977.92
  5228.3  952.86  5264.6  950.16  5279.8  942.89  5299.0  952.44  5338.1  952.86
#Mann=3,-1,0
  4647.1    0.15       0  4969.5    0.05       0  5030.5    0.15       0
Bank Sta=4969.5,5030.5
XS Rating Curve= 0
Exp/Cntr=0.3,0.1

Type RM Length L Ch R = 1,90000,500,500,500
BEGIN DESCRIPTION:
Chauga River 180.0
END DESCRIPTION:
XS GIS Cut Line= 3
      1342311.14      1067701.98      1342106.03      1067620.25
      1341765.85      1067563.39
#Sta/Elev= 30
  4779.2  968.56  4798.5  966.59  4823.9  960.40  4862.1  942.67  4862.2  944.87
  4897.5  933.17  4911.9  923.29  4923.8  918.54  4948.8  900.36  4949.5  899.50
  4949.8  890.73  4951.7  893.88  4957.5  894.46  4968.8  888.74  4969.5  878.39
  4970.0  877.39  5030.5  878.39  5031.6  880.70  5041.2  880.63  5045.2  894.01
  5047.7  915.58  5048.5  881.97  5048.9  878.39  5058.9  887.12  5111.1  897.14
  5120.9  917.05  5146.0  901.32  5168.8  904.90  5288.1  913.77  5344.9  913.19
#Mann=3,-1,0
  4779.2    0.15       0  4969.5    0.05       0  5030.5    0.15       0
Bank Sta=4969.5,5030.5
XS Rating Curve= 0
Exp/Cntr=0.3,0.1

Type RM Length L Ch R = 1,89500,500,500,500
BEGIN DESCRIPTION:
Chauga River 179.0
END DESCRIPTION:
XS GIS Cut Line= 3
      1342398.47      1067518.19      1342343.11      1067188.10
      1342238.80      1066807.22
#Sta/Elev= 30
  4665.3  936.55  4698.6  929.17  4709.4  942.23  4712.3  926.14  4797.9  908.66
  4801.2  899.65  4810.5  906.20  4920.2  882.93  4937.0  889.89  4969.5  876.80
  4970.0  875.80  5030.5  876.80  5054.0  888.04  5062.7  876.80  5072.6  904.72
  5073.6  920.32  5075.6  917.19  5085.4  933.83  5096.8  888.68  5098.8  920.14
  5125.2  978.86  5137.4  994.91  5166.8 1007.59  5207.2 1035.95  5251.6 1055.91
  5259.3 1081.32  5259.9 1066.90  5266.2 1060.81  5356.9 1082.07  5394.9 1080.00
#Mann=3,-1,0
  4665.3    0.15       0  4969.5    0.05       0  5030.5    0.15       0
Bank Sta=4969.5,5030.5
XS Rating Curve= 0
Exp/Cntr=0.3,0.1

Type RM Length L Ch R = 1,89000,500,500,500
BEGIN DESCRIPTION:
Chauga River 178.0
END DESCRIPTION:
XS GIS Cut Line= 3
      1342377.40      1067586.28      1342659.06      1067488.96
      1343097.39      1067417.58
#Sta/Elev= 30
  4702.0  948.31  4729.5  942.52  4735.6  961.08  4748.4  937.53  4861.3  905.62
  4863.4  896.57  4876.4  901.46  4922.2  889.14  4926.3  880.84  4941.2  887.00
  4969.5  876.80  4970.0  875.80  5030.5  876.80  5053.3  885.32  5062.2  876.80
  5063.4  891.34  5075.3  900.62  5079.0  902.18  5081.0  890.76  5083.2  913.55
  5152.4  960.34  5176.9  964.57  5190.2  956.00  5242.6  994.75  5278.4 1010.94
  5349.6 1033.45  5375.2 1033.69  5385.3 1056.31  5394.1 1040.39  5444.1 1055.12
#Mann=3,-1,0
  4702.0    0.15       0  4969.5    0.05       0  5030.5    0.15       0
Bank Sta=4969.5,5030.5
XS Rating Curve= 0
Exp/Cntr=0.3,0.1

Type RM Length L Ch R = 1,88500,500,500,500
BEGIN DESCRIPTION:
Chauga River 177.0
END DESCRIPTION:
XS GIS Cut Line= 3
      1342256.87      1067902.59      1342526.48      1067965.28
      1342799.17      1068026.12
#Sta/Elev= 30
  4723.2  990.23  4733.4  987.13  4762.9  959.73  4810.2  932.67  4834.2  913.72
  4862.2  897.21  4868.5  910.15  4871.7  911.31  4872.8  915.89  4873.0  910.56
  4875.0  888.92  4876.9  884.31  4877.5  886.43  4910.4  882.70  4926.8  878.46
  4928.3  874.32  4929.3  876.67  4969.5  874.32  4970.0  873.32  5030.5  874.32
  5068.0  881.23  5074.5  888.20  5076.6  904.73  5077.2  911.83  5094.6  905.20
  5103.6  906.90  5121.1  916.68  5150.3  917.59  5235.9  934.73  5279.4  939.83
#Mann=3,-1,0
  4723.2    0.15       0  4969.5    0.05       0  5030.5    0.15       0
Bank Sta=4969.5,5030.5
XS Rating Curve= 0
Exp/Cntr=0.3,0.1

Type RM Length L Ch R = 1,88000,500,500,500
BEGIN DESCRIPTION:
Chauga River 176.0
END DESCRIPTION:
XS GIS Cut Line= 3
      1342503.92      1068685.82      1342676.56      1068324.22
      1342937.71      1067836.31
#Sta/Elev= 30
  4599.3  947.70  4705.5  960.42  4707.1  965.41  4709.7  959.52  4723.0  989.08
  4726.9  957.01  4741.4  952.61  4784.5  941.16  4786.1  949.13  4786.5  941.93
  4855.9  946.24  4886.2  940.98  4916.9  912.47  4927.9  891.98  4936.9  883.76
  4969.5  870.50  4970.0  869.50  5030.5  870.50  5041.0  870.65  5041.6  878.34
  5051.3  882.82  5058.2  882.59  5058.7  877.45  5058.9  883.02  5080.5  899.83
  5117.0  898.28  5185.2  923.67  5353.5  944.56  5466.2  950.37  5553.4  965.80
#Mann=3,-1,0
  4599.3    0.15       0  4969.5    0.05       0  5030.5    0.15       0
Bank Sta=4969.5,5030.5
XS Rating Curve= 0
Exp/Cntr=0.3,0.1

Type RM Length L Ch R = 1,87500,500,500,500
BEGIN DESCRIPTION:
Chauga River 175.0
END DESCRIPTION:
XS GIS Cut Line= 3
      1343317.27      1068622.56      1343150.30      1068272.88
      1342970.86      1067869.49
#Sta/Elev= 30
  4612.5 1002.88  4640.6 1013.46  4670.0 1015.64  4690.9 1013.23  4821.0  981.26
  4846.0  969.87  4863.0  958.24  4902.3  922.33  4967.0  874.08  4969.5  869.29
  4970.0  868.29  5030.5  869.29  5051.1  878.65  5054.3  870.65  5057.7  877.57
  5068.8  883.11  5069.6  880.97  5072.5  893.25  5073.3  900.87  5084.5  883.52
  5155.9  896.45  5198.0  913.17  5221.1  918.67  5265.4  924.71  5281.8  924.44
  5302.4  908.17  5310.1  928.65  5388.7  942.31  5430.0  952.45  5441.5  959.10
#Mann=3,-1,0
  4612.5    0.15       0  4969.5    0.05       0  5030.5    0.15       0
Bank Sta=4969.5,5030.5
XS Rating Curve= 0
Exp/Cntr=0.3,0.1

Type RM Length L Ch R = 1,87000,500,500,500
BEGIN DESCRIPTION:
Chauga River 174.0
END DESCRIPTION:
XS GIS Cut Line= 3
      1343924.98      1068424.98      1343590.82      1068036.53
      1343386.58      1067736.92
#Sta/Elev= 30
  4487.6 1005.54  4503.2 1003.19  4621.0  964.09  4705.1  947.67  4775.9  927.85
  4922.9  881.06  4930.5  890.64  4931.9  884.35  4950.5  872.54  4969.3  868.10
  4969.8  867.10  5030.7  868.10  5047.1  869.88  5073.6  881.27  5078.2  892.91
  5079.8  900.87  5085.8  894.57  5109.1  883.51  5162.5  916.88  5170.2  932.56
  5185.3  931.39  5200.7  938.20  5211.9  949.87  5262.6  966.92  5318.3  977.89
  5347.6  995.25  5354.6 1019.51  5356.4 1017.26  5357.9  999.62  5362.6 1008.84
#Mann=3,-1,0
  4487.6    0.15       0  4969.3    0.05       0  5030.7    0.15       0
Bank Sta=4969.3,5030.7
XS Rating Curve= 0
Exp/Cntr=0.3,0.1

Type RM Length L Ch R = 1,86500,500,500,500
BEGIN DESCRIPTION:
Chauga River 173.0
END DESCRIPTION:
XS GIS Cut Line= 3
      1344359.57      1068218.87      1343995.62      1067746.27
      1343702.87      1067541.09
#Sta/Elev= 30
  4403.5 1017.12  4428.9  999.58  4432.8 1004.33  4442.5 1004.96  4508.5  990.40
  4606.7  976.20  4699.6  944.14  4748.7  924.09  4771.6  908.98  4790.4  908.36
  4881.0  887.03  4941.2  881.56  4969.3  866.36  4969.8  865.36  5030.7  866.36
  5065.7  877.87  5069.2  866.68  5072.4  877.00  5107.0  885.79  5120.9  884.89
  5128.0  901.35  5132.7  898.92  5135.2  884.75  5165.5  885.36  5167.4  890.23
  5187.8  897.44  5261.7  945.14  5276.1  946.33  5283.8  951.62  5357.5  956.23
#Mann=3,-1,0
  4403.5    0.15       0  4969.3    0.05       0  5030.7    0.15       0
Bank Sta=4969.3,5030.7
XS Rating Curve= 0
Exp/Cntr=0.3,0.1

Type RM Length L Ch R = 1,86000,500,500,500
BEGIN DESCRIPTION:
Chauga River 172.0
END DESCRIPTION:
XS GIS Cut Line= 3
      1344459.02      1067409.16      1344169.29      1067289.67
      1343606.47      1067183.21
#Sta/Elev= 30
  4686.6  993.56  4743.6  972.61  4791.0  964.83  4830.2  951.01  4871.7  927.89
  4912.1  899.43  4934.1  879.85  4937.3  878.20  4944.3  879.47  4946.5  873.81
  4969.3  864.82  4969.8  863.82  5030.7  864.82  5038.8  865.27  5045.7  871.68
  5059.1  868.56  5059.5  866.68  5067.8  873.39  5083.9  873.72  5085.0  875.80
  5102.6  880.14  5134.9  892.20  5196.5  900.35  5249.1  912.01  5389.4  927.69
  5399.1  924.99  5424.0  933.37  5427.0  931.20  5496.8  957.47  5572.8  979.14
#Mann=3,-1,0
  4686.6    0.15       0  4969.3    0.05       0  5030.7    0.15       0
Bank Sta=4969.3,5030.7
XS Rating Curve= 0
Exp/Cntr=0.3,0.1

Type RM Length L Ch R = 1,85500,370,370,370
BEGIN DESCRIPTION:
Chauga River 171.0
END DESCRIPTION:
XS GIS Cut Line= 3
      1344724.12      1067101.89      1344401.82      1066847.66
      1343856.49      1066619.87
#Sta/Elev= 30
  4589.5 1016.63  4647.9 1000.35  4728.5  964.27  4770.9  955.87  4876.8  920.87
  4915.1  901.56  4952.5  869.88  4955.8  864.13  4960.3  866.56  4969.3  863.70
  4969.8  862.70  5030.7  863.70  5040.6  864.13  5058.1  871.80  5115.4  880.14
  5221.7  887.54  5222.0  896.22  5224.8  901.80  5233.4  888.03  5289.5  900.89
  5306.0  902.43  5307.4  899.25  5328.1  909.19  5354.2  913.46  5390.2  926.35
  5403.1  952.68  5405.9  928.18  5406.4  926.71  5484.9  968.15  5591.0 1014.57
#Mann=3,-1,0
  4589.5    0.15       0  4969.3    0.05       0  5030.7    0.15       0
Bank Sta=4969.3,5030.7
XS Rating Curve= 0
Exp/Cntr=0.3,0.1

Type RM Length L Ch R = 1,85130,759,759,759
BEGIN DESCRIPTION:
Chauga River 170.0
END DESCRIPTION:
XS GIS Cut Line= 3
      1344847.61      1066767.48      1344576.56      1066521.68
      1344125.04      1066275.02
#Sta/Elev= 30
  4634.1  938.69  4661.9  941.13  4740.5  924.73  4881.0  885.55  4910.5  882.23
  4924.2  873.09  4947.0  872.83  4969.3  861.14  4969.8  860.14  5030.7  861.14
  5073.2  871.81  5074.0  869.97  5074.1  861.49  5074.7  871.02  5102.9  872.67
  5108.7  879.87  5119.4  872.00  5125.7  890.93  5134.5  896.85  5203.4  933.00
  5216.6  933.12  5225.7  962.03  5231.7  943.83  5263.6  954.47  5280.4  954.81
  5283.1  960.10  5307.4  969.96  5377.9  984.46  5480.6  980.27  5514.5  971.77
#Mann=3,-1,0
  4634.1    0.15       0  4969.3    0.05       0  5030.7    0.15       0
Bank Sta=4969.3,5030.7
XS Rating Curve= 0
Exp/Cntr=0.3,0.1

Type RM Length L Ch R = 1,84371,371,371,371
BEGIN DESCRIPTION:
Chauga River 169.0
END DESCRIPTION:
XS GIS Cut Line= 3
      1345534.47      1066402.98      1345084.61      1066018.46
      1344669.88      1065640.82
#Sta/Elev= 30
  4408.2 1034.26  4553.1 1002.18  4583.1 1006.70  4613.5  993.63  4628.2  996.88
  4667.3  977.52  4702.5  974.98  4762.8  947.43  4785.3  923.44  4894.7  875.39
  4919.0  910.60  4925.8  930.44  4929.0  901.58  4929.3  890.18  4930.5  869.28
  4969.1  861.09  4969.6  860.09  5030.9  861.09  5044.3  875.87  5050.4  862.36
  5080.8  886.93  5090.8  907.12  5131.0  891.91  5150.3  899.13  5259.7  878.67
  5276.2  889.30  5290.2  889.67  5332.5  916.74  5399.9  941.56  5560.9  973.35
#Mann=3,-1,0
  4408.2    0.15       0  4969.1    0.05       0  5030.9    0.15       0
Bank Sta=4969.1,5030.9
XS Rating Curve= 0
Exp/Cntr=0.3,0.1

Type RM Length L Ch R = 1,84000,500,500,500
BEGIN DESCRIPTION:
Chauga River 168.0
END DESCRIPTION:
XS GIS Cut Line= 3
      1345663.96      1065767.34      1345224.25      1065695.12
      1344736.18      1065661.91
#Sta/Elev= 30
  4554.4  982.34  4579.8  989.24  4657.1  992.98  4765.8  973.85  4798.9  958.57
  4816.3  957.68  4855.2  938.12  4876.5  922.16  4882.9  896.39  4883.0  908.61
  4885.1  919.11  4897.1  917.96  4922.3  898.77  4929.4  874.37  4950.1  855.48
  4969.1  855.48  4969.6  854.48  5030.9  855.48  5046.0  881.47  5051.3  869.46
  5056.5  867.15  5146.6  893.51  5156.8  892.96  5165.5  882.33  5173.3  888.61
  5197.3  892.75  5238.0  884.51  5287.4  886.09  5407.6  942.66  5489.2  961.21
#Mann=3,-1,0
  4554.4    0.15       0  4969.1    0.05       0  5030.9    0.15       0
Bank Sta=4969.1,5030.9
XS Rating Curve= 0
Exp/Cntr=0.3,0.1

Type RM Length L Ch R = 1,83500,500,500,500
BEGIN DESCRIPTION:
Chauga River 167.0
END DESCRIPTION:
XS GIS Cut Line= 3
      1345597.70      1065152.80      1345182.74      1065201.43
      1344802.42      1065216.06
#Sta/Elev= 30
  4582.2  985.41  4611.9  972.59  4620.1  963.97  4677.1  940.12  4682.5  933.50
  4714.5  926.90  4715.7  920.78  4721.3  912.52  4743.8  907.26  4757.6  894.80
  4777.3  894.50  4792.3  881.83  4912.5  873.41  4919.2  863.41  4942.4  862.40
  4969.1  852.36  4969.6  851.36  5030.9  852.36  5045.0  852.38  5053.4  886.93
  5058.4  878.64  5070.9  878.95  5106.6  931.23  5111.1  941.71  5112.7  936.23
  5119.6  940.23  5122.0  927.92  5203.5  960.45  5270.9  973.29  5380.6 1007.64
#Mann=3,-1,0
  4582.2    0.15       0  4969.1    0.05       0  5030.9    0.15       0
Bank Sta=4969.1,5030.9
XS Rating Curve= 0
Exp/Cntr=0.3,0.1

Type RM Length L Ch R = 1,83000,500,500,500
BEGIN DESCRIPTION:
Chauga River 166.0
END DESCRIPTION:
XS GIS Cut Line= 3
      1345700.18      1064661.76      1345338.98      1064755.62
      1344968.16      1064908.77
#Sta/Elev= 30
  4626.8 1013.48  4754.7  967.34  4839.7  950.51  4871.6  931.55  4879.8  863.33
  4881.4  881.54  4894.2  917.00  4905.1  875.88  4905.7  859.59  4909.7  899.49
  4913.9  899.11  4931.3  857.78  4947.0  835.19  4954.6  844.40  4969.1  835.19
  4969.6  834.19  5030.9  835.19  5047.8  842.55  5128.3  838.60  5130.0  864.26
  5135.3  839.27  5154.7  845.73  5163.7  859.79  5164.3  876.04  5166.3  863.92
  5172.3  853.76  5209.8  887.64  5287.4  924.77  5342.7  931.83  5401.2  926.22
#Mann=3,-1,0
  4626.8    0.15       0  4969.1    0.05       0  5030.9    0.15       0
Bank Sta=4969.1,5030.9
XS Rating Curve= 0
Exp/Cntr=0.3,0.1

Type RM Length L Ch R = 1,82500,500,500,500
BEGIN DESCRIPTION:
Chauga River 165.0
END DESCRIPTION:
XS GIS Cut Line= 3
      1345666.97      1064405.69      1345200.54      1064280.66
      1344841.57      1064212.90
#Sta/Elev= 30
  4517.1  980.30  4576.4  976.42  4584.6  989.56  4596.4  969.96  4754.3  904.13
  4804.9  890.91  4824.1  865.53  4841.6  853.67  4900.8  846.47  4902.0  861.04
  4902.6  847.73  4904.7  845.60  4905.6  860.62  4905.7  848.22  4906.5  846.17
  4969.1  832.89  4969.6  831.89  5030.9  832.89  5040.1  836.20  5040.9  849.47
  5043.3  862.87  5047.4  843.37  5084.7  868.05  5085.9  855.31  5086.0  844.93
  5087.5  872.38  5090.8  881.70  5191.6  948.74  5294.3  993.85  5365.3  997.25
#Mann=3,-1,0
  4517.1    0.15       0  4969.1    0.05       0  5030.9    0.15       0
Bank Sta=4969.1,5030.9
XS Rating Curve= 0
Exp/Cntr=0.3,0.1

Type RM Length L Ch R = 1,82000,500,500,500
BEGIN DESCRIPTION:
Chauga River 164.0
END DESCRIPTION:
XS GIS Cut Line= 3
      1345862.79      1063808.03      1345337.83      1063801.24
      1345085.63      1063820.07
#Sta/Elev= 30
  4475.0 1076.03  4566.3 1032.98  4622.5 1017.95  4637.4 1004.89  4693.0 1002.35
  4737.3  967.80  4764.1  963.03  4788.9  935.82  4830.5  915.45  4854.1  890.88
  4883.2  876.50  4889.8  847.17  4899.3  861.30  4933.0  839.60  4936.9  830.39
  4969.1  830.39  4969.6  829.39  5030.9  830.39  5037.7  835.10  5043.0  863.04
  5056.5  838.27  5086.3  842.41  5104.6  851.79  5106.8  863.50  5110.7  844.47
  5111.1  852.09  5113.8  857.13  5122.2  863.43  5188.2  901.68  5252.9  919.66
#Mann=3,-1,0
  4475.0    0.15       0  4969.1    0.05       0  5030.9    0.15       0
Bank Sta=4969.1,5030.9
XS Rating Curve= 0
Exp/Cntr=0.3,0.1

Type RM Length L Ch R = 1,81500,500,500,500
BEGIN DESCRIPTION:
Chauga River 163.0
END DESCRIPTION:
XS GIS Cut Line= 3
      1345178.99      1063142.28      1345103.95      1063451.81
      1345019.33      1063844.19
#Sta/Elev= 30
  4681.5  987.12  4696.5  983.00  4698.0  992.35  4718.8  997.67  4791.5 1002.33
  4837.7 1014.20  4861.7  953.79  4888.3  919.20  4898.2  886.84  4902.7  850.17
  4903.1  874.74  4909.6  895.39  4933.4  852.53  4942.0  842.46  4955.9  838.02
  4964.6  824.16  4964.9  833.00  4965.5  834.14  4969.1  824.02  4969.6  823.02
  5030.9  824.02  5038.7  824.02  5073.2  844.34  5097.5  843.81  5103.6  852.45
  5116.6  851.24  5178.1  872.57  5249.1  888.60  5328.9  894.60  5401.4  922.81
#Mann=3,-1,0
  4681.5    0.15       0  4969.1    0.05       0  5030.9    0.15       0
Bank Sta=4969.1,5030.9
XS Rating Curve= 0
Exp/Cntr=0.3,0.1

Type RM Length L Ch R = 1,81000,436,436,436
BEGIN DESCRIPTION:
Chauga River 162.0
END DESCRIPTION:
XS GIS Cut Line= 3
      1344672.89      1063392.27      1344687.09      1063674.52
      1344690.97      1064088.20
#Sta/Elev= 30
  4717.4  955.05  4812.0  931.71  4830.2  922.19  4843.5  908.23  4869.7  894.99
  4874.0  841.97  4875.0  835.97  4899.8  846.24  4913.8  858.58  4955.4  824.64
  4956.3  822.06  4959.5  827.60  4966.0  826.69  4969.1  822.06  4969.6  821.06
  5030.9  822.06  5039.2  828.78  5045.0  822.12  5049.5  831.05  5056.2  837.80
  5069.7  842.05  5073.4  839.28  5152.6  868.69  5228.1  885.17  5248.5  883.17
  5255.6  895.47  5334.9  942.07  5356.7  951.39  5398.8  959.08  5413.7  963.86
#Mann=3,-1,0
  4717.4    0.15       0  4969.1    0.05       0  5030.9    0.15       0
Bank Sta=4969.1,5030.9
XS Rating Curve= 0
Exp/Cntr=0.3,0.1

Type RM Length L Ch R = 1,80564,564,564,564
BEGIN DESCRIPTION:
Chauga River 161.0
END DESCRIPTION:
XS GIS Cut Line= 3
      1344588.56      1063392.30      1344290.40      1063560.63
      1344019.21      1063838.13
#Sta/Elev= 30
  4657.6  925.51  4677.5  915.48  4729.2  897.00  4783.5  869.68  4840.5  861.74
  4892.3  844.77  4915.9  842.51  4925.0  853.96  4936.5  841.08  4945.1  842.73
  4965.1  836.64  4968.0  828.71  4969.0  820.59  4969.5  819.59  5031.0  820.59
  5038.7  820.59  5042.9  835.55  5047.1  842.90  5059.9  856.82  5067.5  857.60
  5111.7  906.98  5155.2  932.87  5160.9  927.07  5161.1  930.01  5163.0  935.17
  5193.2  943.91  5244.8  946.98  5286.6  966.13  5331.0  968.64  5388.0  959.22
#Mann=3,-1,0
  4657.6    0.15       0  4969.0    0.05       0  5031.0    0.15       0
Bank Sta=4969,5031
XS Rating Curve= 0
Exp/Cntr=0.3,0.1

Type RM Length L Ch R = 1,80000,500,500,500
BEGIN DESCRIPTION:
Chauga River 160.0
END DESCRIPTION:
XS GIS Cut Line= 3
      1344672.89      1063060.93      1344310.43      1063012.37
      1343856.48      1062934.40
#Sta/Elev= 30
  4634.3  966.68  4693.4  945.16  4760.7  911.28  4800.4  895.54  4810.7  888.56
  4886.3  868.90  4895.9  868.55  4917.5  900.67  4927.3  850.91  4932.8  845.80
  4940.2  834.22  4948.1  837.01  4965.7  827.96  4969.0  818.63  4969.5  817.63
  5031.0  818.63  5043.3  827.14  5061.4  832.13  5105.6  838.45  5109.8  836.92
  5203.2  871.24  5229.6  883.69  5294.0  902.31  5333.8  928.13  5344.5  932.05
  5395.1  963.11  5442.2  981.20  5446.1  979.32  5448.6  982.40  5460.6  982.83
#Mann=3,-1,0
  4634.3    0.15       0  4969.0    0.05       0  5031.0    0.15       0
Bank Sta=4969,5031
XS Rating Curve= 0
Exp/Cntr=0.3,0.1

Type RM Length L Ch R = 1,79500,500,500,500
BEGIN DESCRIPTION:
Chauga River 159.0
END DESCRIPTION:
XS GIS Cut Line= 3
      1344901.81      1062751.23      1344433.94      1062528.00
      1344022.20      1062428.91
#Sta/Elev= 30
  4481.6  931.87  4652.8  894.30  4808.7  846.85  4891.9  844.15  4952.6  835.24
  4968.1  824.16  4969.0  817.00  4969.5  816.00  5031.0  817.00  5048.2  822.32
  5076.6  850.30  5077.3  839.44  5078.9  836.41  5081.9  854.47  5090.7  861.60
  5091.4  853.42  5092.4  863.36  5109.7  875.41  5119.4  892.64  5140.3  901.55
  5168.1  921.99  5183.2  925.80  5215.3  918.78  5276.1  882.66  5276.7  888.12
  5278.6  890.50  5297.7  903.38  5358.9  938.31  5389.6  952.10  5423.5  960.13
#Mann=3,-1,0
  4481.6    0.15       0  4969.0    0.05       0  5031.0    0.15       0
Bank Sta=4969,5031
XS Rating Curve= 0
Exp/Cntr=0.3,0.1

Type RM Length L Ch R = 1,79000,500,500,500
BEGIN DESCRIPTION:
Chauga River 158.0
END DESCRIPTION:
XS GIS Cut Line= 3
      1345019.34      1062359.63      1344681.97      1062101.65
      1344260.23      1061989.10
#Sta/Elev= 30
  4575.3  979.83  4613.0  968.83  4615.2  961.51  4628.8  965.54  4759.4  909.08
  4793.4  890.55  4809.8  870.07  4816.2  854.75  4818.3  866.68  4823.4  867.78
  4855.2  837.98  4947.8  837.35  4964.6  830.85  4969.0  816.77  4969.5  815.77
  5031.0  816.77  5098.0  855.55  5112.6  857.96  5133.8  856.87  5145.5  828.03
  5153.9  851.51  5170.8  839.27  5178.4  848.41  5236.3  845.36  5279.7  866.15
  5289.6  899.47  5292.3  875.05  5298.8  883.69  5304.6  871.00  5436.5  900.70
#Mann=3,-1,0
  4575.3    0.15       0  4969.0    0.05       0  5031.0    0.15       0
Bank Sta=4969,5031
XS Rating Curve= 0
Exp/Cntr=0.3,0.1

Type RM Length L Ch R = 1,78500,500,500,500
BEGIN DESCRIPTION:
Chauga River 157.0
END DESCRIPTION:
XS GIS Cut Line= 3
      1345338.67      1061868.60      1344973.71      1061699.81
      1344474.96      1061524.99
#Sta/Elev= 30
  4597.9  959.97  4652.3  950.03  4760.1  974.15  4791.7  963.99  4804.2  984.07
  4831.0  957.65  4874.4  936.21  4957.6  864.38  4964.5  847.67  4965.4  857.21
  4968.4  848.13  4969.0  816.77  4969.5  815.77  5031.0  816.77  5036.9  826.62
  5050.5  832.44  5127.9  832.26  5163.9  837.63  5165.4  844.28  5167.3  838.26
  5256.0  839.05  5273.4  856.17  5285.7  841.23  5310.1  847.33  5384.5  887.90
  5389.2  897.89  5413.3  905.83  5457.5  950.19  5499.6  977.89  5528.5  982.89
#Mann=3,-1,0
  4597.9    0.15       0  4969.0    0.05       0  5031.0    0.15       0
Bank Sta=4969,5031
XS Rating Curve= 0
Exp/Cntr=0.3,0.1

Type RM Length L Ch R = 1,78000,500,500,500
BEGIN DESCRIPTION:
Chauga River 156.0
END DESCRIPTION:
XS GIS Cut Line= 3
      1345597.74      1061326.35      1345152.33      1061232.92
      1344675.93      1061097.40
#Sta/Elev= 30
  4544.9  919.76  4559.6  913.86  4578.1  910.62  4593.5  902.82  4611.2  901.73
  4659.8  890.05  4670.1  884.98  4690.9  884.02  4825.0  847.20  4857.3  843.45
  4893.9  824.41  4908.8  829.31  4933.4  830.12  4958.3  826.32  4969.0  816.86
  4969.5  815.86  5031.0  816.86  5054.1  831.55  5069.4  834.39  5105.2  830.31
  5130.0  830.30  5148.1  833.63  5191.9  857.61  5198.6  864.09  5214.3  868.35
  5269.5  897.14  5377.2  961.80  5413.4  979.97  5460.3  995.36  5495.3  999.35
#Mann=3,-1,0
  4544.9    0.15       0  4969.0    0.05       0  5031.0    0.15       0
Bank Sta=4969,5031
XS Rating Curve= 0
Exp/Cntr=0.3,0.1

Type RM Length L Ch R = 1,77500,436,436,436
BEGIN DESCRIPTION:
Chauga River 155.0
END DESCRIPTION:
XS GIS Cut Line= 3
      1345751.36      1061022.08      1345429.30      1060820.95
      1345145.87      1060651.55
#Sta/Elev= 30
  4620.3  898.76  4663.8  883.42  4668.8  894.51  4674.3  901.36  4680.1  884.49
  4687.1  890.94  4690.8  886.98  4693.9  873.22  4744.4  856.17  4804.5  843.73
  4871.5  839.74  4935.1  830.33  4961.0  821.00  4963.5  822.63  4968.9  816.18
  4969.4  815.18  5031.1  816.18  5034.1  816.25  5046.6  828.99  5060.1  835.63
  5060.4  829.43  5064.8  835.55  5066.2  839.75  5121.4  868.46  5228.6  916.60
  5249.9  924.34  5286.6  932.90  5316.2  934.09  5319.4  936.01  5330.2  932.51
#Mann=3,-1,0
  4620.3    0.15       0  4968.9    0.05       0  5031.1    0.15       0
Bank Sta=4968.9,5031.1
XS Rating Curve= 0
Exp/Cntr=0.3,0.1

Type RM Length L Ch R = 1,77064,564,564,564
BEGIN DESCRIPTION:
Chauga River 154.0
END DESCRIPTION:
XS GIS Cut Line= 3
      1346075.02      1060875.02      1345727.89      1060504.80
      1345474.25      1060346.10
#Sta/Elev= 30
  4492.5  954.54  4515.5  955.02  4517.2  971.27  4523.2  962.59  4529.2  970.90
  4536.5  953.22  4560.0  950.33  4612.6  933.93  4636.1  925.80  4665.1  911.78
  4697.2  900.79  4822.8  867.84  4898.2  836.65  4935.7  832.59  4968.4  819.68
  4968.9  815.40  4969.4  814.40  5031.1  815.40  5033.3  824.37  5034.5  815.40
  5034.6  823.92  5037.0  826.99  5051.4  830.46  5082.1  830.46  5084.1  833.47
  5110.5  842.01  5149.5  859.26  5184.1  869.47  5246.8  873.46  5299.2  870.67
#Mann=3,-1,0
  4492.5    0.15       0  4968.9    0.05       0  5031.1    0.15       0
Bank Sta=4968.9,5031.1
XS Rating Curve= 0
Exp/Cntr=0.3,0.1

Type RM Length L Ch R = 1,76500,354,354,354
BEGIN DESCRIPTION:
Chauga River 153.0
END DESCRIPTION:
XS GIS Cut Line= 3
      1346396.02      1060096.04      1345938.20      1059996.13
      1345447.13      1059942.41
#Sta/Elev= 30
  4531.4  971.15  4609.3  967.45  4658.2  962.79  4764.4  942.88  4792.2  935.33
  4856.1  911.82  4862.9  907.06  4874.5  894.48  4882.7  891.28  4911.5  868.75
  4920.2  892.89  4920.7  898.78  4921.0  895.14  4929.7  853.38  4946.8  833.91
  4957.4  826.78  4968.9  813.81  4969.4  812.81  5031.1  813.81  5032.8  822.82
  5040.9  826.61  5055.9  828.82  5074.3  822.77  5117.9  825.46  5197.7  841.98
  5221.8  843.14  5319.4  857.31  5346.6  859.39  5386.0  867.79  5494.0  895.08
#Mann=3,-1,0
  4531.4    0.15       0  4968.9    0.05       0  5031.1    0.15       0
Bank Sta=4968.9,5031.1
XS Rating Curve= 0
Exp/Cntr=0.3,0.1

Type RM Length L Ch R = 1,76146,351,351,351
BEGIN DESCRIPTION:
Chauga River 152.0
END DESCRIPTION:
XS GIS Cut Line= 3
      1346269.48      1059692.37      1345977.48      1059645.09
      1345480.27      1059617.06
#Sta/Elev= 30
  4704.2  905.35  4724.0  909.58  4745.8  909.45  4748.3  906.06  4752.8  910.30
  4761.6  909.51  4836.5  891.55  4854.2  883.55  4886.5  861.95  4911.1  837.93
  4915.3  829.27  4917.9  835.87  4930.1  829.85  4962.9  825.40  4968.9  812.14
  4969.4  811.14  5031.1  812.14  5037.5  815.09  5041.1  812.22  5044.2  821.32
  5050.6  826.85  5065.0  830.78  5132.0  835.65  5180.3  846.59  5259.9  857.25
  5340.8  875.93  5342.3  873.01  5352.0  878.97  5443.0  897.09  5498.0  903.25
#Mann=3,-1,0
  4704.2    0.15       0  4968.9    0.05       0  5031.1    0.15       0
Bank Sta=4968.9,5031.1
XS Rating Curve= 0
Exp/Cntr=0.3,0.1

Type RM Length L Ch R = 1,75795,667,667,667
BEGIN DESCRIPTION:
Chauga River 151.0
END DESCRIPTION:
XS GIS Cut Line= 3
      1346465.32      1059321.84      1346028.18      1059297.82
      1345471.18      1059312.80
#Sta/Elev= 30
  4562.2  907.58  4675.5  888.10  4731.3  874.67  4843.0  841.79  4901.0  834.68
  4915.1  829.85  4954.0  825.07  4965.1  820.04  4968.9  812.22  4969.4  811.22
  5031.1  812.22  5041.8  819.30  5043.7  812.22  5050.3  827.33  5056.5  824.46
  5068.8  830.83  5113.1  831.32  5232.3  838.52  5252.9  837.90  5256.8  840.90
  5281.3  846.37  5295.4  852.18  5356.3  864.11  5391.1  866.16  5412.7  872.04
  5445.9  876.50  5461.1  880.87  5469.6  885.51  5516.6  894.08  5557.2  897.97
#Mann=3,-1,0
  4562.2    0.15       0  4968.9    0.05       0  5031.1    0.15       0
Bank Sta=4968.9,5031.1
XS Rating Curve= 0
Exp/Cntr=0.3,0.1

Type RM Length L Ch R = 1,75128,628,628,628
BEGIN DESCRIPTION:
Chauga River 150.0
END DESCRIPTION:
XS GIS Cut Line= 3
      1346486.42      1058697.65      1346091.89      1058633.59
      1345543.55      1058592.22
#Sta/Elev= 30
  4600.3  878.11  4699.8  893.85  4747.6  893.68  4786.2  887.48  4811.3  880.55
  4905.9  837.87  4909.5  832.89  4918.5  832.92  4955.2  822.22  4957.9  824.60
  4966.2  820.60  4968.9  811.43  4969.4  810.43  5031.1  811.43  5041.5  821.78
  5042.2  811.43  5045.0  818.79  5050.5  824.83  5087.6  827.49  5093.5  824.69
  5096.5  829.54  5115.1  824.79  5127.4  814.39  5137.5  820.93  5139.6  819.83
  5144.4  826.02  5146.3  822.78  5178.6  823.28  5286.9  829.85  5549.9  938.57
#Mann=3,-1,0
  4600.3    0.15       0  4968.9    0.05       0  5031.1    0.15       0
Bank Sta=4968.9,5031.1
XS Rating Curve= 0
Exp/Cntr=0.3,0.1

Type RM Length L Ch R = 1,74500,500,500,500
BEGIN DESCRIPTION:
Chauga River 149.0
END DESCRIPTION:
XS GIS Cut Line= 3
      1346528.60      1058045.75      1346172.29      1058011.00
      1345767.52      1057992.51
#Sta/Elev= 30
  4642.0  879.76  4697.8  873.19  4748.7  863.34  4777.7  853.22  4812.3  834.37
  4817.1  830.45  4818.0  832.21  4841.7  828.88  4912.3  829.58  4949.8  825.62
  4955.7  822.81  4961.4  822.49  4968.9  810.66  4969.4  809.66  5031.1  810.66
  5035.5  812.32  5035.8  810.72  5045.2  820.94  5051.0  824.33  5054.2  822.76
  5086.2  829.23  5166.2  822.94  5262.0  824.12  5266.7  826.86  5282.4  822.77
  5303.5  830.89  5310.8  831.03  5339.1  839.36  5381.4  858.68  5405.2  866.65
#Mann=3,-1,0
  4642.0    0.15       0  4968.9    0.05       0  5031.1    0.15       0
Bank Sta=4968.9,5031.1
XS Rating Curve= 0
Exp/Cntr=0.3,0.1

Type RM Length L Ch R = 1,74000,500,500,500
BEGIN DESCRIPTION:
Chauga River 148.0
END DESCRIPTION:
XS GIS Cut Line= 3
      1346865.98      1057937.30      1346285.55      1057529.27
      1346076.71      1057422.16
#Sta/Elev= 30
  4290.5  904.21  4375.0  891.07  4488.7  888.82  4490.8  886.30  4546.4  877.72
  4633.8  856.70  4772.2  833.66  4958.7  821.51  4968.3  817.80  4968.9  809.67
  4969.4  808.67  5031.1  809.67  5033.5  815.81  5035.5  809.67  5038.2  811.80
  5041.5  819.33  5041.9  815.73  5042.2  821.15  5046.3  829.87  5056.3  837.06
  5059.2  858.03  5062.5  865.58  5068.0  872.13  5068.4  862.69  5076.2  864.03
  5100.8  888.68  5110.1  891.35  5142.7  916.99  5187.0  933.35  5234.7  938.24
#Mann=3,-1,0
  4290.5    0.15       0  4968.9    0.05       0  5031.1    0.15       0
Bank Sta=4968.9,5031.1
XS Rating Curve= 0
Exp/Cntr=0.3,0.1

Type RM Length L Ch R = 1,73500,500,500,500
BEGIN DESCRIPTION:
Chauga River 147.0
END DESCRIPTION:
XS GIS Cut Line= 3
      1346965.44      1056952.20      1346480.44      1057093.28
      1346010.46      1057322.74
#Sta/Elev= 30
  4494.9  935.41  4684.0  911.78  4701.3  907.58  4825.2  901.24  4849.0  897.22
  4851.5  893.68  4873.9  882.68  4892.7  865.63  4904.7  859.64  4917.5  843.43
  4945.7  824.11  4948.3  819.33  4954.0  821.30  4956.3  818.71  4957.4  809.24
  4958.1  811.40  4968.6  809.24  4969.1  808.24  5031.4  809.24  5041.9  817.43
  5110.1  821.33  5136.1  832.06  5191.9  844.42  5262.2  855.12  5289.7  861.66
  5306.0  868.95  5327.7  871.45  5377.4  887.26  5474.3  905.56  5523.0  911.69
#Mann=3,-1,0
  4494.9    0.15       0  4968.6    0.05       0  5031.4    0.15       0
Bank Sta=4968.6,5031.4
XS Rating Curve= 0
Exp/Cntr=0.3,0.1

Type RM Length L Ch R = 1,73000,428,428,428
BEGIN DESCRIPTION:
Chauga River 146.0
END DESCRIPTION:
XS GIS Cut Line= 3
      1346477.40      1056500.32      1346104.05      1056786.32
      1345733.26      1057069.73
#Sta/Elev= 30
  4529.7  909.89  4577.0  905.22  4666.4  925.08  4714.7  919.89  4749.2  910.74
  4801.0  885.27  4810.2  873.74  4826.9  861.27  4838.5  862.38  4879.0  850.43
  4887.3  831.66  4888.4  839.36  4894.2  829.51  4927.4  827.45  4938.0  820.61
  4946.1  820.21  4956.4  809.24  4959.8  814.06  4968.6  809.24  4969.1  808.24
  5031.4  809.24  5036.5  815.83  5043.0  818.07  5121.0  821.16  5168.2  827.82
  5175.4  834.90  5195.7  841.30  5303.4  867.23  5307.7  871.16  5466.7  920.45
#Mann=3,-1,0
  4529.7    0.15       0  4968.6    0.05       0  5031.4    0.15       0
Bank Sta=4968.6,5031.4
XS Rating Curve= 0
Exp/Cntr=0.3,0.1

Type RM Length L Ch R = 1,72572,199,199,199
BEGIN DESCRIPTION:
Chauga River 145.0
END DESCRIPTION:
XS GIS Cut Line= 3
      1346041.43      1056302.50      1345786.76      1056498.73
      1345397.84      1056912.70
#Sta/Elev= 30
  4678.5  874.80  4774.5  862.85  4776.4  860.84  4783.1  860.54  4805.6  852.60
  4822.0  843.54  4856.7  842.97  4868.0  835.93  4890.6  826.51  4898.0  819.80
  4899.0  821.57  4915.3  820.38  4922.6  815.21  4934.6  812.52  4935.4  809.24
  4942.6  811.12  4968.6  809.24  4969.1  808.24  5031.4  809.24  5033.4  816.96
  5105.0  820.51  5131.4  828.65  5165.0  828.42  5177.9  833.23  5179.8  832.23
  5213.8  839.67  5248.7  853.12  5385.9  868.71  5480.7  889.87  5568.0  901.52
#Mann=3,-1,0
  4678.5    0.15       0  4968.6    0.05       0  5031.4    0.15       0
Bank Sta=4968.6,5031.4
XS Rating Curve= 0
Exp/Cntr=0.3,0.1

Type RM Length L Ch R = 1,72373,373,373,373
BEGIN DESCRIPTION:
Chauga River 144.5
END DESCRIPTION:
XS GIS Cut Line= 3
      1345953.41      1056244.82      1345685.71      1056333.46
      1345246.11      1056451.24
#Sta/Elev= 30
  4718.0  856.71  4783.4  848.50  4823.5  835.47  4848.6  823.72  4863.2  821.75
  4871.6  817.47  4900.7  815.16  4924.9  808.26  4968.6  807.91  4969.1  806.91
  5031.4  807.91  5052.0  809.47  5112.2  808.04  5121.7  812.07  5157.6  818.17
  5171.0  827.96  5178.6  827.73  5184.9  831.17  5238.8  830.39  5244.8  833.83
  5246.9  836.97  5276.4  846.94  5313.6  854.59  5339.4  852.44  5377.1  864.43
  5399.4  866.41  5414.3  860.97  5414.8  858.74  5419.4  865.07  5455.1  859.13
#Mann=3,-1,0
  4718.0    0.15       0  4968.6    0.05       0  5031.4    0.15       0
Bank Sta=4968.6,5031.4
XS Rating Curve= 0
Exp/Cntr=0.3,0.1

Type RM Length L Ch R = 1,72000,397,397,397
BEGIN DESCRIPTION:
Chauga River 144.0
END DESCRIPTION:
XS GIS Cut Line= 3
      1346100.84      1056234.06      1345807.82      1056010.12
      1345531.47      1055792.42
#Sta/Elev= 30
  4631.2  874.19  4636.0  871.14  4698.0  870.30  4723.7  863.06  4726.3  865.67
  4735.9  858.32  4785.2  845.41  4830.2  824.50  4892.1  807.80  4926.9  803.95
  4939.4  798.03  4968.6  798.03  4969.1  797.03  5031.4  798.03  5033.8  801.00
  5035.0  798.30  5041.7  809.45  5044.2  810.25  5044.7  804.10  5057.1  817.35
  5073.3  844.89  5113.6  867.70  5154.2  879.99  5177.0  882.40  5184.4  895.58
  5184.5  889.98  5194.5  886.61  5200.9  892.89  5251.2  902.71  5351.8  906.51
#Mann=3,-1,0
  4631.2    0.15       0  4968.6    0.05       0  5031.4    0.15       0
Bank Sta=4968.6,5031.4
XS Rating Curve= 0
Exp/Cntr=0.3,0.1

Type RM Length L Ch R = 1,71603,497,497,497
BEGIN DESCRIPTION:
Chauga River 143.0
END DESCRIPTION:
XS GIS Cut Line= 3
      1346374.91      1055727.94      1345965.51      1055662.46
      1345546.52      1055616.48
#Sta/Elev= 30
  4585.4  883.77  4653.2  867.64  4675.8  868.34  4745.9  842.81  4764.1  843.26
  4780.3  837.60  4809.2  816.18  4830.5  815.55  4854.6  805.34  4959.0  802.45
  4965.0  800.73  4968.6  797.16  4969.1  796.16  5031.4  797.16  5047.0  797.16
  5052.7  804.99  5064.8  812.67  5078.2  816.70  5122.2  837.36  5144.6  845.64
  5180.5  852.38  5254.0  857.78  5323.5  867.79  5358.1  873.41  5361.9  877.62
  5362.0  874.29  5363.0  874.24  5377.1  878.11  5395.0  877.77  5421.5  886.11
#Mann=3,-1,0
  4585.4    0.15       0  4968.6    0.05       0  5031.4    0.15       0
Bank Sta=4968.6,5031.4
XS Rating Curve= 0
Exp/Cntr=0.3,0.1

Type RM Length L Ch R = 1,71106,606,606,606
BEGIN DESCRIPTION:
Chauga River 142.0
END DESCRIPTION:
XS GIS Cut Line= 3
      1346468.29      1055414.62      1346162.70      1055208.16
      1345874.83      1055050.11
#Sta/Elev= 30
  4631.2  838.66  4702.4  838.15  4766.6  848.60  4821.3  848.80  4855.8  837.93
  4928.0  803.47  4968.6  793.99  4969.1  792.99  5031.4  793.99  5060.7  795.30
  5068.5  800.92  5071.9  807.36  5073.6  814.22  5082.4  805.83  5095.9  824.13
  5098.3  821.86  5106.5  839.85  5109.6  833.36  5113.9  842.20  5114.7  848.96
  5128.2  850.00  5128.3  840.31  5132.4  854.05  5157.2  857.90  5187.8  875.73
  5216.2  883.80  5223.1  880.85  5225.3  884.16  5253.3  883.28  5328.4  900.78
#Mann=3,-1,0
  4631.2    0.15       0  4968.6    0.05       0  5031.4    0.15       0
Bank Sta=4968.6,5031.4
XS Rating Curve= 0
Exp/Cntr=0.3,0.1

Type RM Length L Ch R = 1,70500,371,371,371
BEGIN DESCRIPTION:
Chauga River 141.0
END DESCRIPTION:
XS GIS Cut Line= 3
      1346896.14      1054860.36      1346500.86      1054709.76
      1346073.74      1054528.99
#Sta/Elev= 30
  4577.0  930.83  4705.6  889.38  4711.8  885.70  4712.1  879.68  4714.5  886.12
  4739.7  870.61  4785.2  858.85  4798.5  847.09  4827.8  839.01  4829.4  842.83
  4861.4  821.35  4905.2  806.27  4908.2  799.82  4968.6  792.28  4969.1  791.28
  5031.4  792.28  5060.2  796.57  5060.3  800.75  5067.8  804.35  5068.5  812.22
  5072.2  805.64  5151.9  859.83  5166.4  875.42  5187.3  880.17  5201.6  890.34
  5203.4  908.25  5223.2  904.38  5277.8  919.10  5341.8  921.98  5463.8  907.87
#Mann=3,-1,0
  4577.0    0.15       0  4968.6    0.05       0  5031.4    0.15       0
Bank Sta=4968.6,5031.4
XS Rating Curve= 0
Exp/Cntr=0.3,0.1

Type RM Length L Ch R = 1,70129,629,629,629
BEGIN DESCRIPTION:
Chauga River 140.0
END DESCRIPTION:
XS GIS Cut Line= 3
      1347122.18      1054499.92      1346669.71      1054381.15
      1346247.82      1054184.18
#Sta/Elev= 30
  4532.2  934.09  4550.9  934.71  4557.8  929.57  4580.4  927.17  4608.5  916.88
  4643.0  896.38  4672.4  891.65  4675.8  894.90  4704.8  884.45  4715.3  889.16
  4738.0  883.26  4795.7  837.48  4820.2  815.17  4823.3  807.39  4824.6  811.09
  4829.7  804.50  4963.4  789.03  4967.1  787.52  4968.6  781.93  4969.1  780.93
  5031.4  781.93  5081.5  782.28  5098.6  796.88  5113.4  817.98  5161.7  846.67
  5228.0  854.59  5323.4  836.75  5419.9  873.75  5429.8  881.30  5465.6  890.88
#Mann=3,-1,0
  4532.2    0.15       0  4968.6    0.05       0  5031.4    0.15       0
Bank Sta=4968.6,5031.4
XS Rating Curve= 0
Exp/Cntr=0.3,0.1

Type RM Length L Ch R = 1,69500,500,500,500
BEGIN DESCRIPTION:
Chauga River 139.0
END DESCRIPTION:
XS GIS Cut Line= 3
      1347311.86      1053938.54      1346928.69      1053835.04
      1346459.32      1053718.62
#Sta/Elev= 30
  4603.1  898.31  4626.2  899.83  4705.3  885.27  4787.1  867.37  4794.4  864.51
  4796.1  860.71  4803.3  862.55  4816.5  853.30  4831.8  854.94  4848.5  852.31
  4899.2  832.31  4934.4  812.09  4943.8  809.80  4958.1  789.36  4959.5  791.54
  4968.6  779.19  4969.1  778.19  5031.4  779.19  5061.1  783.69  5061.5  779.22
  5062.0  781.61  5069.5  786.83  5109.3  794.48  5185.0  813.86  5229.1  835.48
  5254.5  851.75  5286.7  855.68  5296.4  866.85  5318.9  874.96  5483.6  911.65
#Mann=3,-1,0
  4603.1    0.15       0  4968.6    0.05       0  5031.4    0.15       0
Bank Sta=4968.6,5031.4
XS Rating Curve= 0
Exp/Cntr=0.3,0.1

Type RM Length L Ch R = 1,69000,500,500,500
BEGIN DESCRIPTION:
Chauga River 138.0
END DESCRIPTION:
XS GIS Cut Line= 3
      1347637.18      1053580.04      1347094.79      1053367.62
      1346902.17      1053296.88
#Sta/Elev= 30
  4417.5  845.09  4504.7  848.82  4621.3  831.27  4657.8  801.03  4663.6  798.88
  4665.3  810.29  4665.6  799.01  4705.3  790.20  4712.9  783.98  4769.1  802.05
  4864.5  791.65  4924.1  791.37  4956.1  786.05  4968.6  774.67  4969.1  773.67
  5031.4  774.67  5044.0  798.68  5052.1  774.67  5058.6  800.89  5058.9  778.88
  5059.0  787.07  5064.2  798.63  5065.3  809.96  5065.6  797.47  5066.7  784.80
  5078.0  822.02  5091.7  833.79  5111.6  843.06  5120.2  853.08  5205.2  855.33
#Mann=3,-1,0
  4417.5    0.15       0  4968.6    0.05       0  5031.4    0.15       0
Bank Sta=4968.6,5031.4
XS Rating Curve= 0
Exp/Cntr=0.3,0.1

Type RM Length L Ch R = 1,68500,500,500,500
BEGIN DESCRIPTION:
Chauga River 137.0
END DESCRIPTION:
XS GIS Cut Line= 3
      1347721.50      1052700.42      1347341.46      1052955.12
      1346932.24      1053275.80
#Sta/Elev= 30
  4542.5  964.19  4638.4  946.50  4691.4  951.27  4767.1  947.77  4768.1  942.88
  4772.1  940.59  4808.8  932.86  4835.7  916.40  4868.8  846.24  4896.7  820.36
  4935.7  802.15  4940.0  787.45  4940.5  796.78  4961.5  774.30  4965.0  783.31
  4968.5  774.30  4969.0  773.30  5031.5  774.30  5049.9  784.61  5130.4  789.85
  5143.8  794.99  5143.9  790.93  5163.6  805.46  5211.5  818.93  5256.7  822.87
  5321.6  841.13  5392.3  853.44  5455.4  852.94  5486.4  844.41  5519.9  851.02
#Mann=3,-1,0
  4542.5    0.15       0  4968.5    0.05       0  5031.5    0.15       0
Bank Sta=4968.5,5031.5
XS Rating Curve= 0
Exp/Cntr=0.3,0.1

Type RM Length L Ch R = 1,68000,500,500,500
BEGIN DESCRIPTION:
Chauga River 136.0
END DESCRIPTION:
XS GIS Cut Line= 3
      1346902.14      1052555.76      1346874.00      1052870.51
      1346835.86      1053278.83
#Sta/Elev= 30
  4684.0  940.66  4715.5  937.08  4727.1  945.92  4729.3  933.05  4795.3  899.87
  4824.1  889.86  4867.6  858.73  4901.3  855.92  4914.0  850.40  4925.9  843.10
  4940.6  823.02  4942.1  823.89  4946.8  797.09  4947.0  779.41  4949.8  779.84
  4953.0  804.24  4953.9  804.51  4958.1  786.72  4959.9  774.43  4962.9  777.21
  4968.5  774.25  4969.0  773.25  5031.5  774.25  5040.5  783.31  5079.0  790.76
  5219.5  804.98  5233.7  808.45  5245.8  816.41  5286.8  818.95  5410.1  860.67
#Mann=3,-1,0
  4684.0    0.15       0  4968.5    0.05       0  5031.5    0.15       0
Bank Sta=4968.5,5031.5
XS Rating Curve= 0
Exp/Cntr=0.3,0.1

Type RM Length L Ch R = 1,67500,500,500,500
BEGIN DESCRIPTION:
Chauga River 135.0
END DESCRIPTION:
XS GIS Cut Line= 3
      1346393.02      1052603.99      1346380.23      1052946.76
      1346411.10      1053447.51
#Sta/Elev= 30
  4657.0  870.81  4702.6  865.24  4728.2  858.48  4802.9  844.55  4827.4  837.47
  4880.1  816.85  4909.4  797.35  4922.8  791.84  4930.7  784.80  4946.2  785.89
  4954.2  783.58  4955.7  785.26  4965.2  781.72  4968.5  772.41  4969.0  771.41
  5031.5  772.41  5036.0  772.41  5045.4  783.95  5085.6  789.73  5121.7  797.66
  5150.8  805.58  5243.0  840.41  5252.7  843.26  5270.1  842.59  5284.9  849.87
  5295.9  859.54  5359.4  881.23  5386.4  886.00  5452.0  890.49  5501.7  902.23
#Mann=3,-1,0
  4657.0    0.15       0  4968.5    0.05       0  5031.5    0.15       0
Bank Sta=4968.5,5031.5
XS Rating Curve= 0
Exp/Cntr=0.3,0.1

Type RM Length L Ch R = 1,67000,500,500,500
BEGIN DESCRIPTION:
Chauga River 134.0
END DESCRIPTION:
XS GIS Cut Line= 3
      1346444.22      1052508.81      1346047.42      1052643.68
      1345570.58      1052864.29
#Sta/Elev= 30
  4580.9  870.52  4677.2  863.04  4724.6  851.99  4741.1  843.99  4768.8  845.12
  4794.9  841.05  4835.8  826.98  4883.5  799.02  4922.0  794.56  4968.0  780.47
  4968.5  772.41  4969.0  771.41  5031.5  772.41  5036.7  772.41  5042.0  777.21
  5057.9  782.53  5089.8  788.05  5103.1  794.93  5116.3  795.14  5147.1  806.50
  5170.3  805.82  5172.3  806.85  5172.8  812.37  5174.0  814.08  5317.7  867.65
  5366.9  875.38  5393.5  876.88  5420.3  874.72  5430.3  877.71  5525.4  883.98
#Mann=3,-1,0
  4580.9    0.15       0  4968.5    0.05       0  5031.5    0.15       0
Bank Sta=4968.5,5031.5
XS Rating Curve= 0
Exp/Cntr=0.3,0.1

Type RM Length L Ch R = 1,66500,500,500,500
BEGIN DESCRIPTION:
Chauga River 133.0
END DESCRIPTION:
XS GIS Cut Line= 3
      1346456.30      1052141.28      1346004.86      1052148.78
      1345552.55      1052068.98
#Sta/Elev= 30
  4548.5  882.02  4707.7  862.69  4800.5  829.34  4844.1  807.72  4900.4  790.99
  4940.6  785.84  4944.6  782.48  4955.6  781.06  4961.2  777.12  4963.5  774.16
  4963.9  770.39  4964.0  773.36  4967.0  774.34  4968.5  770.39  4969.0  769.39
  5031.5  770.39  5044.0  770.52  5058.5  781.20  5080.9  787.06  5107.3  797.76
  5136.2  816.40  5162.0  826.65  5174.9  835.91  5178.0  835.34  5211.6  849.41
  5248.5  858.34  5296.1  864.00  5399.9  854.45  5437.6  854.59  5459.3  857.47
#Mann=3,-1,0
  4548.5    0.15       0  4968.5    0.05       0  5031.5    0.15       0
Bank Sta=4968.5,5031.5
XS Rating Curve= 0
Exp/Cntr=0.3,0.1

Type RM Length L Ch R = 1,66000,401,401,401
BEGIN DESCRIPTION:
Chauga River 132.0
END DESCRIPTION:
XS GIS Cut Line= 3
      1346516.07      1051886.07      1346079.35      1051657.32
      1345643.91      1051503.54
#Sta/Elev= 30
  4507.0  848.46  4546.3  852.00  4592.5  845.51  4624.9  834.76  4693.8  804.01
  4708.8  804.51  4755.4  798.67  4783.1  798.97  4869.9  786.94  4946.1  785.37
  4958.4  781.98  4963.8  776.00  4966.2  777.12  4967.7  768.62  4968.2  767.62
  5032.3  768.62  5036.1  769.43  5036.6  773.38  5047.3  778.35  5078.0  784.62
  5107.0  795.71  5118.8  797.93  5127.1  804.83  5133.7  802.07  5148.5  803.51
  5200.7  799.56  5317.5  823.83  5356.6  824.78  5358.3  822.55  5461.8  836.32
#Mann=3,-1,0
  4507.0    0.15       0  4967.7    0.05       0  5032.3    0.15       0
Bank Sta=4967.7,5032.3
XS Rating Curve= 0
Exp/Cntr=0.3,0.1

Type RM Length L Ch R = 1,65599,492,492,492
BEGIN DESCRIPTION:
Chauga River 131.0
END DESCRIPTION:
XS GIS Cut Line= 3
      1346783.83      1051745.81      1346279.42      1051312.14
      1346067.17      1051209.21
#Sta/Elev= 30
  4334.8  827.29  4432.4  817.74  4468.1  803.55  4488.2  791.80  4520.2  787.39
  4570.2  794.46  4594.6  793.61  4596.7  790.84  4663.6  791.27  4703.0  799.55
  4704.1  796.16  4705.6  799.94  4818.1  787.97  4854.9  790.08  4933.0  781.75
  4948.8  784.15  4966.7  773.64  4967.7  767.76  4968.2  766.76  5032.3  767.76
  5035.4  774.48  5050.2  780.80  5101.6  779.92  5136.2  800.77  5168.6  815.51
  5206.8  818.24  5215.3  825.54  5216.5  821.77  5225.2  818.83  5235.9  818.83
#Mann=3,-1,0
  4334.8    0.15       0  4967.7    0.05       0  5032.3    0.15       0
Bank Sta=4967.7,5032.3
XS Rating Curve= 0
Exp/Cntr=0.3,0.1

Type RM Length L Ch R = 1,65107,607,607,607
BEGIN DESCRIPTION:
Chauga River 130.0
END DESCRIPTION:
XS GIS Cut Line= 3
      1346839.93      1051859.55      1346663.84      1051027.38
      1346638.45      1050775.65
#Sta/Elev= 30
  4149.4  849.43  4452.7  805.29  4541.5  783.09  4558.5  782.04  4574.5  794.50
  4575.8  786.49  4575.9  792.50  4576.4  794.02  4591.0  796.66  4630.4  797.11
  4656.2  790.06  4684.0  793.27  4685.4  786.95  4695.5  795.73  4728.8  797.43
  4795.9  788.32  4893.6  788.23  4898.2  780.97  4948.9  778.47  4967.7  766.27
  4968.2  765.27  5032.3  766.27  5044.6  778.73  5050.6  772.61  5075.3  808.93
  5096.9  826.14  5150.6  847.86  5173.7  870.33  5198.7  878.88  5253.0  913.87
#Mann=3,-1,0
  4149.4    0.15       0  4967.7    0.05       0  5032.3    0.15       0
Bank Sta=4967.7,5032.3
XS Rating Curve= 0
Exp/Cntr=0.3,0.1

Type RM Length L Ch R = 1,64500,608,608,608
BEGIN DESCRIPTION:
Chauga River 129.0
END DESCRIPTION:
XS GIS Cut Line= 3
      1346931.72      1051893.73      1347181.43      1051301.20
      1347230.11      1051083.48
#Sta/Elev= 30
  4357.0  861.95  4469.1  821.02  4541.6  800.50  4569.7  799.76  4589.6  791.43
  4624.0  806.12  4712.5  810.22  4791.7  799.14  4824.1  789.25  4824.6  791.76
  4858.1  789.96  4879.7  784.76  4940.0  780.90  4960.9  775.42  4966.1  772.12
  4967.7  765.60  4968.2  764.60  5032.3  765.60  5035.1  765.60  5041.9  780.38
  5045.7  771.14  5045.8  774.10  5049.2  782.24  5053.1  784.92  5053.7  778.57
  5054.2  796.09  5070.3  806.34  5109.3  811.89  5177.6  845.80  5223.1  850.19
#Mann=3,-1,0
  4357.0    0.15       0  4967.7    0.05       0  5032.3    0.15       0
Bank Sta=4967.7,5032.3
XS Rating Curve= 0
Exp/Cntr=0.3,0.1
