HEC-RAS study Chauga River.prj: Chauga River Limited Detail Study

--- Chauga River.g01 (geometry) --- (continued)

Type RM Length L Ch R = 1,63892,392,392,392
BEGIN DESCRIPTION:
Chauga River 128.0
END DESCRIPTION:
XS GIS Cut Line= 3
      1347737.61      1052017.16      1347716.89      1051570.84
      1347683.03      1051356.40
#Sta/Elev= 30
  4553.2  863.78  4590.7  869.03  4690.0  857.23  4835.7  788.51  4855.1  783.03
  4906.0  783.05  4930.2  779.57  4956.8  772.58  4967.7  764.19  4968.2  763.19
  5032.3  764.19  5033.6  782.28  5034.7  782.86  5035.7  778.85  5037.8  764.19
  5045.5  786.41  5049.9  788.40  5057.5  781.79  5059.2  790.69  5062.9  794.38
  5063.4  793.01  5063.7  779.52  5064.3  790.90  5066.7  795.69  5078.4  798.62
  5102.4  811.93  5122.6  813.24  5134.9  822.44  5163.2  835.23  5217.1  842.52
#Mann=3,-1,0
  4553.2    0.15       0  4967.7    0.05       0  5032.3    0.15       0
Bank Sta=4967.7,5032.3
XS Rating Curve= 0
Exp/Cntr=0.3,0.1

Type RM Length L Ch R = 1,63500,500,500,500
BEGIN DESCRIPTION:
Chauga River 127.0
END DESCRIPTION:
XS GIS Cut Line= 3
      1348391.98      1051539.99      1348054.61      1051424.46
      1347711.06      1051315.56
#Sta/Elev= 30
  4643.4  874.63  4668.4  876.14  4720.7  875.67  4737.6  877.10  4782.9  885.20
  4795.2  886.12  4810.9  886.11  4831.7  881.83  4837.7  878.01  4840.8  881.38
  4842.6  880.47  4859.3  860.63  4898.9  836.44  4911.2  832.55  4915.8  826.30
  4950.1  795.36  4957.0  763.70  4964.6  766.86  4967.7  763.70  4968.2  762.70
  5031.8  762.70  5032.3  763.70  5047.6  775.82  5058.9  778.10  5192.3  784.99
  5233.0  789.54  5252.4  795.53  5292.6  813.61  5311.9  820.69  5360.4  835.79
#Mann=3,-1,0
  4643.4    0.15       0  4967.7    0.05       0  5032.3    0.15       0
Bank Sta=4967.7,5032.3
XS Rating Curve= 0
Exp/Cntr=0.3,0.1

Type RM Length L Ch R = 1,63000,500,500,500
BEGIN DESCRIPTION:
Chauga River 126.0
END DESCRIPTION:
XS GIS Cut Line= 3
      1348315.45      1050822.37      1347999.90      1050945.70
      1347626.90      1051110.54
#Sta/Elev= 30
  4661.2  858.53  4715.8  849.99  4734.3  844.52  4768.9  838.37  4842.3  829.07
  4859.4  828.74  4885.9  821.78  4891.8  822.56  4898.7  817.58  4937.2  802.79
  4939.0  804.42  4954.1  786.36  4965.6  775.45  4967.7  762.20  4968.2  761.20
  5032.3  762.20  5040.6  770.03  5047.7  773.99  5047.9  772.43  5049.2  774.16
  5123.4  782.23  5172.0  781.74  5210.6  786.14  5212.1  783.86  5214.4  786.29
  5229.7  790.96  5263.0  806.86  5289.7  816.84  5359.2  836.80  5407.8  847.48
#Mann=3,-1,0
  4661.2    0.15       0  4967.7    0.05       0  5032.3    0.15       0
Bank Sta=4967.7,5032.3
XS Rating Curve= 0
Exp/Cntr=0.3,0.1

Type RM Length L Ch R = 1,62500,354,354,354
BEGIN DESCRIPTION:
Chauga River 125.0
END DESCRIPTION:
XS GIS Cut Line= 3
      1348221.08      1050458.19      1347788.86      1050498.53
      1347356.58      1050567.85
#Sta/Elev= 30
  4565.9  851.08  4646.3  832.44  4711.3  812.20  4740.4  801.41  4775.8  792.55
  4800.6  787.73  4856.8  780.99  4863.2  778.83  4863.8  777.10  4864.7  779.23
  4867.4  779.80  4886.1  771.11  4940.8  770.38  4951.6  767.01  4951.7  762.72
  4953.1  765.34  4967.7  760.54  4968.2  759.54  5032.3  760.54  5048.2  771.20
  5076.8  777.28  5088.4  774.69  5129.8  776.78  5131.3  774.85  5150.6  782.62
  5226.6  820.59  5262.0  831.67  5308.8  836.89  5384.6  841.79  5437.8  847.16
#Mann=3,-1,0
  4565.9    0.15       0  4967.7    0.05       0  5032.3    0.15       0
Bank Sta=4967.7,5032.3
XS Rating Curve= 0
Exp/Cntr=0.3,0.1

Type RM Length L Ch R = 1,62146,403,403,403
BEGIN DESCRIPTION:
Chauga River 124.0
END DESCRIPTION:
XS GIS Cut Line= 3
      1348157.35      1050363.05      1347712.22      1050170.23
      1347377.03      1050077.44
#Sta/Elev= 30
  4514.9  832.80  4635.2  791.23  4663.8  783.33  4667.3  786.84  4670.2  781.96
  4820.2  774.29  4829.9  768.74  4843.8  767.54  4961.3  772.97  4963.9  770.61
  4967.6  757.43  4968.1  756.43  5032.4  757.43  5050.8  766.48  5056.9  773.55
  5057.5  777.00  5058.0  773.30  5059.2  777.18  5060.6  773.39  5061.6  785.95
  5073.4  798.96  5092.6  805.01  5099.4  813.03  5106.4  813.46  5151.5  841.21
  5178.6  853.23  5226.8  864.26  5247.1  880.67  5251.2  870.99  5347.8  885.98
#Mann=3,-1,0
  4514.9    0.15       0  4967.6    0.05       0  5032.4    0.15       0
Bank Sta=4967.6,5032.4
XS Rating Curve= 0
Exp/Cntr=0.3,0.1

Type RM Length L Ch R = 1,61743,500,500,500
BEGIN DESCRIPTION:
Chauga River 123.0
END DESCRIPTION:
XS GIS Cut Line= 3
      1348310.38      1050312.56      1348033.85      1049995.11
      1347756.99      1049761.72
#Sta/Elev= 30
  4579.0  851.37  4625.6  847.54  4635.3  843.65  4641.2  846.36  4674.4  835.22
  4702.0  832.03  4755.9  812.67  4795.0  789.72  4797.5  793.90  4799.2  788.91
  4806.6  786.04  4860.3  778.03  4933.2  774.91  4945.2  772.12  4952.7  773.86
  4960.9  757.43  4967.6  757.43  4968.1  756.43  5032.4  757.43  5037.5  757.51
  5044.9  765.25  5060.4  770.83  5063.4  774.19  5126.8  785.76  5170.8  797.82
  5257.7  833.98  5324.4  855.44  5328.2  858.59  5332.0  856.55  5362.1  860.71
#Mann=3,-1,0
  4579.0    0.15       0  4967.6    0.05       0  5032.4    0.15       0
Bank Sta=4967.6,5032.4
XS Rating Curve= 0
Exp/Cntr=0.3,0.1

Type RM Length L Ch R = 1,61243,696,696,696
BEGIN DESCRIPTION:
Chauga River 122.0
END DESCRIPTION:
XS GIS Cut Line= 3
      1348366.49      1050316.92      1348385.07      1049668.39
      1348374.14      1049261.13
#Sta/Elev= 30
  4351.2  845.00  4400.9  838.37  4466.9  819.14  4479.4  811.53  4501.8  812.70
  4518.0  808.10  4544.9  804.35  4553.3  805.67  4572.1  801.73  4600.5  794.13
  4643.0  776.69  4647.9  776.64  4648.0  778.51  4648.5  775.90  4965.5  768.76
  4967.6  757.43  4968.1  756.43  5032.4  757.43  5050.3  757.43  5076.9  775.04
  5089.0  770.22  5089.1  773.85  5116.5  791.91  5124.2  794.70  5142.4  797.99
  5196.2  814.77  5236.3  822.90  5297.4  830.82  5367.6  827.95  5407.4  821.82
#Mann=3,-1,0
  4351.2    0.15       0  4967.6    0.05       0  5032.4    0.15       0
Bank Sta=4967.6,5032.4
XS Rating Curve= 0
Exp/Cntr=0.3,0.1

Type RM Length L Ch R = 1,60547,547,547,547
BEGIN DESCRIPTION:
Chauga River 121.0
END DESCRIPTION:
XS GIS Cut Line= 3
      1348348.60      1050471.72      1348761.44      1050229.60
      1349144.30      1049989.72
#Sta/Elev= 30
  4521.4  862.38  4560.7  856.17  4578.7  849.15  4585.9  850.20  4637.1  834.41
  4708.9  818.16  4715.7  812.95  4737.0  812.59  4788.5  795.16  4832.1  783.55
  4947.3  768.99  4948.3  770.57  4961.9  764.66  4966.4  758.45  4967.1  759.97
  4967.6  757.00  4968.1  756.00  5032.4  757.00  5033.8  764.64  5035.1  757.21
  5038.3  763.81  5042.2  767.47  5049.3  768.20  5056.9  772.67  5082.8  775.89
  5147.8  801.64  5240.8  805.22  5326.9  819.04  5390.1  814.43  5451.8  825.90
#Mann=3,-1,0
  4521.4    0.15       0  4967.6    0.05       0  5032.4    0.15       0
Bank Sta=4967.6,5032.4
XS Rating Curve= 0
Exp/Cntr=0.3,0.1

Type RM Length L Ch R = 1,60000,412,412,412
BEGIN DESCRIPTION:
Chauga River 120.0
END DESCRIPTION:
XS GIS Cut Line= 3
      1348664.91      1050907.26      1349007.47      1050717.92
      1349358.54      1050483.94
#Sta/Elev= 30
  4608.6  811.99  4676.5  823.29  4720.5  826.64  4720.8  827.89  4722.4  826.52
  4758.7  824.93  4759.7  825.14  4759.9  826.73  4828.4  804.96  4865.7  788.97
  4901.7  770.84  4922.7  766.75  4942.0  767.60  4953.6  765.87  4963.5  761.94
  4967.6  755.37  4968.1  754.37  5032.4  755.37  5040.4  765.30  5046.2  767.94
  5068.8  767.20  5133.0  772.21  5261.0  773.99  5278.8  777.82  5294.1  778.19
  5294.7  776.35  5297.3  779.33  5367.7  804.54  5386.3  808.93  5421.9  813.70
#Mann=3,-1,0
  4608.6    0.15       0  4967.6    0.05       0  5032.4    0.15       0
Bank Sta=4967.6,5032.4
XS Rating Curve= 0
Exp/Cntr=0.3,0.1

Type RM Length L Ch R = 1,59588,588,588,588
BEGIN DESCRIPTION:
Chauga River 119.0
END DESCRIPTION:
XS GIS Cut Line= 3
      1349223.37      1051394.40      1349274.24      1051013.38
      1349389.13      1050430.40
#Sta/Elev= 30
  4615.6  917.34  4706.6  887.30  4749.8  869.24  4788.0  850.09  4804.8  845.86
  4835.3  844.91  4860.3  838.52  4870.3  832.45  4871.9  833.18  4905.0  813.09
  4935.3  781.35  4967.6  754.74  4968.1  753.74  5032.4  754.74  5039.4  758.17
  5039.6  754.74  5040.8  758.16  5046.1  763.55  5050.4  765.21  5077.3  764.78
  5140.4  770.84  5224.4  770.20  5341.0  771.85  5368.7  773.58  5417.1  791.95
  5460.4  804.18  5475.2  805.02  5479.7  807.14  5513.6  811.22  5594.2  816.85
#Mann=3,-1,0
  4615.6    0.15       0  4967.6    0.05       0  5032.4    0.15       0
Bank Sta=4967.6,5032.4
XS Rating Curve= 0
Exp/Cntr=0.3,0.1

Type RM Length L Ch R = 1,59000,450,450,450
BEGIN DESCRIPTION:
Chauga River 118.0
END DESCRIPTION:
XS GIS Cut Line= 3
      1349940.48      1051121.48      1349781.81      1050726.13
      1349631.92      1050376.83
#Sta/Elev= 30
  4574.0  825.99  4659.1  803.90  4701.6  797.82  4713.3  794.07  4787.4  779.83
  4896.7  768.60  4943.4  766.91  4949.3  765.14  4951.2  762.65  4961.9  756.40
  4962.7  754.15  4967.6  754.11  4968.1  753.11  5032.4  754.11  5034.6  762.48
  5038.3  763.70  5039.1  761.91  5039.7  757.72  5043.0  766.01  5048.5  768.19
  5050.9  764.53  5055.6  767.02  5099.2  771.68  5120.3  771.92  5141.9  775.47
  5179.1  793.62  5224.0  811.04  5257.8  819.07  5310.4  825.79  5380.1  828.56
#Mann=3,-1,0
  4574.0    0.15       0  4967.6    0.05       0  5032.4    0.15       0
Bank Sta=4967.6,5032.4
XS Rating Curve= 0
Exp/Cntr=0.3,0.1

Type RM Length L Ch R = 1,58550,550,550,550
BEGIN DESCRIPTION:
Chauga River 117.0
END DESCRIPTION:
XS GIS Cut Line= 3
      1350230.22      1050636.45      1350148.90      1050467.17
      1349997.57      1050227.44
#Sta/Elev= 30
  4812.2  778.69  4827.3  780.59  4869.0  779.42  4937.8  760.71  4942.5  761.80
  4951.0  752.92  4955.3  755.15  4967.6  752.92  4968.1  751.92  5032.4  752.92
  5037.0  762.46  5041.3  764.31  5044.8  763.72  5045.4  759.47  5045.7  762.84
  5048.0  764.66  5085.1  771.13  5097.8  778.43  5101.3  783.78  5118.2  791.43
  5128.3  793.02  5137.3  799.56  5145.3  802.57  5148.2  800.05  5166.9  809.64
  5168.8  803.12  5171.1  807.07  5172.5  813.14  5196.9  822.32  5283.5  828.67
#Mann=3,-1,0
  4812.2    0.15       0  4967.6    0.05       0  5032.4    0.15       0
Bank Sta=4967.6,5032.4
XS Rating Curve= 0
Exp/Cntr=0.3,0.1

Type RM Length L Ch R = 1,58000,500,500,500
BEGIN DESCRIPTION:
Chauga River 116.0
END DESCRIPTION:
XS GIS Cut Line= 3
      1350858.59      1050351.85      1350569.35      1050113.03
      1350170.04      1049864.76
#Sta/Elev= 30
  4624.9  827.10  4665.0  826.71  4747.2  809.79  4759.0  804.98  4762.5  799.86
  4766.0  803.95  4782.6  795.28  4804.1  798.39  4894.9  772.29  4919.4  769.68
  4934.5  761.21  4939.5  763.01  4951.5  758.60  4953.9  752.78  4961.2  754.89
  4967.4  752.21  4967.9  751.21  5032.6  752.21  5032.9  758.94  5035.7  761.24
  5036.2  760.12  5036.7  752.21  5038.5  758.80  5040.7  761.47  5056.5  762.46
  5074.8  768.80  5339.0  775.37  5418.6  820.73  5451.1  833.09  5470.2  835.13
#Mann=3,-1,0
  4624.9    0.15       0  4967.4    0.05       0  5032.6    0.15       0
Bank Sta=4967.4,5032.6
XS Rating Curve= 0
Exp/Cntr=0.3,0.1

Type RM Length L Ch R = 1,57500,500,500,500
BEGIN DESCRIPTION:
Chauga River 115.0
END DESCRIPTION:
XS GIS Cut Line= 3
      1351156.96      1050010.63      1350894.53      1049734.42
      1350379.14      1049416.42
#Sta/Elev= 30
  4619.0  832.31  4676.6  828.02  4703.0  823.33  4712.7  819.12  4754.1  813.35
  4806.5  797.23  4858.7  777.49  4908.0  766.75  4942.9  762.55  4953.3  758.76
  4962.7  759.12  4965.3  752.78  4967.4  752.21  4967.9  751.21  5032.6  752.21
  5037.7  754.18  5038.7  752.21  5042.8  758.90  5057.7  768.09  5059.2  766.62
  5101.5  770.56  5347.8  768.67  5424.5  770.79  5441.2  772.90  5455.4  779.11
  5475.9  782.63  5480.4  786.14  5572.2  823.40  5592.9  827.79  5605.6  828.38
#Mann=3,-1,0
  4619.0    0.15       0  4967.4    0.05       0  5032.6    0.15       0
Bank Sta=4967.4,5032.6
XS Rating Curve= 0
Exp/Cntr=0.3,0.1

Type RM Length L Ch R = 1,57000,682,682,682
BEGIN DESCRIPTION:
Chauga River 114.0
END DESCRIPTION:
XS GIS Cut Line= 3
      1351466.23      1049673.80      1351233.26      1049366.66
      1351014.17      1049112.97
#Sta/Elev= 30
  4614.5  799.04  4620.3  798.90  4621.8  799.96  4639.0  796.83  4711.6  775.92
  4721.2  774.15  4755.6  769.79  4867.6  766.98  4916.0  762.11  4936.2  761.53
  4946.4  760.30  4960.7  752.35  4965.9  753.41  4967.4  752.35  4967.9  751.35
  5032.1  751.35  5032.6  752.35  5036.8  754.55  5041.0  752.51  5041.1  759.39
  5042.1  760.31  5065.0  765.14  5067.6  767.74  5181.8  765.16  5218.5  766.48
  5240.6  775.01  5269.7  790.48  5296.6  801.04  5314.8  806.02  5335.2  805.66
#Mann=3,-1,0
  4614.5    0.15       0  4967.4    0.05       0  5032.6    0.15       0
Bank Sta=4967.4,5032.6
XS Rating Curve= 0
Exp/Cntr=0.3,0.1

Type RM Length L Ch R = 1,56318,376,376,376
BEGIN DESCRIPTION:
Chauga River 113.0
END DESCRIPTION:
XS GIS Cut Line= 3
      1352098.52      1049446.02      1351751.18      1048925.83
      1351519.03      1048696.38
#Sta/Elev= 30
  4374.5  819.02  4471.6  810.71  4531.2  808.80  4557.4  804.08  4623.7  784.28
  4623.8  780.00  4626.3  780.89  4669.0  764.77  4781.4  764.72  4946.5  758.92
  4955.7  756.59  4958.5  751.91  4963.3  754.29  4967.4  749.54  4967.9  748.54
  5032.6  749.54  5033.8  749.54  5035.4  759.15  5036.8  760.47  5045.3  760.08
  5050.3  764.69  5051.8  763.29  5062.0  766.58  5108.2  793.33  5146.5  804.92
  5146.7  802.77  5164.1  807.75  5225.9  816.81  5300.9  820.73  5326.4  827.34
#Mann=3,-1,0
  4374.5    0.15       0  4967.4    0.05       0  5032.6    0.15       0
Bank Sta=4967.4,5032.6
XS Rating Curve= 0
Exp/Cntr=0.3,0.1

Type RM Length L Ch R = 1,55942,442,442,442
BEGIN DESCRIPTION:
Chauga River 112.0
END DESCRIPTION:
XS GIS Cut Line= 3
      1352386.68      1048708.98      1352008.11      1048660.19
      1351703.69      1048631.19
#Sta/Elev= 30
  4618.3  847.16  4638.6  846.10  4696.5  838.36  4749.0  827.77  4800.2  813.71
  4888.9  781.68  4901.8  774.55  4907.8  765.76  4914.4  768.25  4927.0  761.84
  4940.3  759.80  4942.1  758.17  4946.9  749.54  4949.5  753.24  4957.1  753.53
  4961.3  756.18  4966.0  755.58  4967.3  749.54  4967.8  748.54  5032.7  749.54
  5051.4  749.54  5060.2  756.92  5073.5  758.28  5098.8  764.84  5159.1  792.66
  5270.9  836.72  5271.7  838.74  5272.0  837.62  5277.6  838.98  5305.8  847.17
#Mann=3,-1,0
  4618.3    0.15       0  4967.3    0.05       0  5032.7    0.15       0
Bank Sta=4967.3,5032.7
XS Rating Curve= 0
Exp/Cntr=0.3,0.1

Type RM Length L Ch R = 1,55500,500,500,500
BEGIN DESCRIPTION:
Chauga River 111.0
END DESCRIPTION:
XS GIS Cut Line= 3
      1352514.67      1048253.76      1352082.61      1048225.38
      1351668.03      1048197.66
#Sta/Elev= 30
  4567.0  832.52  4594.1  826.12  4636.7  829.18  4678.5  829.24  4708.2  825.38
  4739.8  824.22  4767.4  818.77  4873.4  784.51  4877.0  779.03  4896.7  765.97
  4904.4  744.31  4907.4  755.16  4930.8  746.92  4958.8  750.98  4967.3  744.31
  4967.8  743.31  5032.7  744.31  5036.5  747.42  5049.9  749.59  5076.6  751.25
  5086.3  749.53  5095.1  754.77  5116.9  760.67  5158.2  780.31  5171.9  791.01
  5185.2  793.81  5264.6  828.94  5304.4  842.89  5340.4  852.69  5415.5  865.58
#Mann=3,-1,0
  4567.0    0.15       0  4967.3    0.05       0  5032.7    0.15       0
Bank Sta=4967.3,5032.7
XS Rating Curve= 0
Exp/Cntr=0.3,0.1

Type RM Length L Ch R = 1,55000,500,500,500
BEGIN DESCRIPTION:
Chauga River 110.0
END DESCRIPTION:
XS GIS Cut Line= 3
      1352489.21      1047760.30      1352087.81      1047730.66
      1351647.59      1047722.04
#Sta/Elev= 30
  4597.5  888.09  4641.1  873.30  4642.6  864.39  4643.1  863.85  4653.9  868.97
  4687.1  862.69  4726.1  851.62  4757.2  845.74  4827.9  820.64  4843.6  810.43
  4893.2  788.13  4920.8  766.69  4929.1  763.97  4938.6  740.31  4947.2  744.78
  4962.4  743.60  4967.3  740.31  4967.8  739.31  5032.7  740.31  5039.1  742.42
  5059.2  740.31  5073.3  751.21  5143.8  779.50  5186.5  793.42  5195.5  794.02
  5218.1  800.37  5322.8  804.02  5348.8  806.81  5401.3  816.03  5440.3  818.73
#Mann=3,-1,0
  4597.5    0.15       0  4967.3    0.05       0  5032.7    0.15       0
Bank Sta=4967.3,5032.7
XS Rating Curve= 0
Exp/Cntr=0.3,0.1

Type RM Length L Ch R = 1,54500,500,500,500
BEGIN DESCRIPTION:
Chauga River 109.0
END DESCRIPTION:
XS GIS Cut Line= 3
      1352445.87      1047256.63      1352122.67      1047232.57
      1351713.90      1047185.21
#Sta/Elev= 30
  4675.9  827.29  4795.8  809.08  4800.8  804.73  4806.9  806.78  4840.7  797.89
  4895.3  777.58  4929.6  757.95  4946.2  751.67  4955.5  737.93  4958.0  745.22
  4962.6  745.09  4967.3  737.93  4967.8  736.93  5032.7  737.93  5038.0  747.70
  5045.0  749.25  5110.6  755.97  5162.7  763.39  5172.4  762.95  5175.1  765.27
  5243.6  778.91  5262.8  785.26  5282.2  787.92  5284.8  786.70  5298.4  793.58
  5312.0  798.25  5351.5  808.32  5382.1  813.71  5390.8  810.67  5411.5  812.49
#Mann=3,-1,0
  4675.9    0.15       0  4967.3    0.05       0  5032.7    0.15       0
Bank Sta=4967.3,5032.7
XS Rating Curve= 0
Exp/Cntr=0.3,0.1

Type RM Length L Ch R = 1,54000,500,500,500
BEGIN DESCRIPTION:
Chauga River 108.0
END DESCRIPTION:
XS GIS Cut Line= 3
      1352458.63      1046988.88      1352223.31      1046754.68
      1351989.36      1046506.87
#Sta/Elev= 30
  4668.0  803.11  4751.3  790.33  4824.9  773.65  4833.5  773.38  4835.0  771.37
  4876.0  759.38  4941.9  747.63  4964.6  737.93  4966.2  739.96  4967.3  737.93
  4967.8  736.93  5032.7  737.93  5040.3  737.93  5045.5  743.54  5046.7  746.52
  5063.0  752.00  5083.6  761.90  5103.7  773.54  5107.7  777.28  5108.2  775.68
  5108.3  778.41  5123.7  782.86  5132.9  788.21  5159.9  799.25  5193.7  810.40
  5206.5  813.49  5220.6  810.23  5225.1  817.35  5252.4  822.06  5340.8  824.50
#Mann=3,-1,0
  4668.0    0.15       0  4967.3    0.05       0  5032.7    0.15       0
Bank Sta=4967.3,5032.7
XS Rating Curve= 0
Exp/Cntr=0.3,0.1

Type RM Length L Ch R = 1,53500,500,500,500
BEGIN DESCRIPTION:
Chauga River 107.0
END DESCRIPTION:
XS GIS Cut Line= 3
      1352530.00      1047014.35      1352624.65      1046484.43
      1352642.21      1046177.84
#Sta/Elev= 30
  4461.7  806.56  4526.3  789.58  4552.7  785.18  4606.5  781.13  4692.7  765.23
  4766.9  758.42  4893.3  754.16  4920.9  751.18  4923.3  747.21  4946.2  742.33
  4950.1  737.24  4967.3  736.60  4967.8  735.60  5032.7  736.60  5044.1  741.76
  5053.5  740.85  5057.2  736.60  5059.9  753.01  5060.6  753.65  5098.9  770.34
  5115.5  767.23  5118.1  771.44  5182.3  770.85  5182.6  774.22  5183.4  774.56
  5262.6  802.05  5293.2  807.59  5293.9  807.38  5294.1  804.70  5307.1  810.03
#Mann=3,-1,0
  4461.7    0.15       0  4967.3    0.05       0  5032.7    0.15       0
Bank Sta=4967.3,5032.7
XS Rating Curve= 0
Exp/Cntr=0.3,0.1

Type RM Length L Ch R = 1,53000,500,500,500
BEGIN DESCRIPTION:
Chauga River 106.0
END DESCRIPTION:
XS GIS Cut Line= 3
      1353340.96      1046331.14      1353024.54      1046243.99
      1352639.65      1046137.32
#Sta/Elev= 30
  4671.8  879.96  4765.6  864.36  4801.4  851.54  4827.1  838.00  4854.3  820.40
  4905.8  782.77  4913.2  780.77  4921.5  774.49  4926.9  765.97  4937.7  753.14
  4947.3  738.34  4948.0  734.78  4948.4  737.49  4950.1  738.94  4961.5  733.96
  4967.3  733.81  4967.8  732.81  5032.7  733.81  5035.2  742.34  5043.3  743.94
  5051.9  748.25  5055.8  745.72  5094.2  748.33  5114.1  752.15  5196.3  759.90
  5270.4  783.15  5275.9  786.32  5276.3  784.76  5332.5  801.86  5399.4  814.59
#Mann=3,-1,0
  4671.8    0.15       0  4967.3    0.05       0  5032.7    0.15       0
Bank Sta=4967.3,5032.7
XS Rating Curve= 0
Exp/Cntr=0.3,0.1

Type RM Length L Ch R = 1,52500,593,593,593
BEGIN DESCRIPTION:
Chauga River 105.0
END DESCRIPTION:
XS GIS Cut Line= 3
      1353453.16      1046065.89      1353147.00      1045761.11
      1352884.51      1045566.10
#Sta/Elev= 30
  4568.0  874.48  4664.5  838.54  4670.5  833.04  4708.0  827.85  4770.3  811.52
  4851.7  783.84  4890.4  768.64  4899.5  760.15  4913.5  758.01  4956.2  734.78
  4967.3  734.49  4967.8  733.49  5032.7  734.49  5050.5  739.17  5053.1  734.78
  5062.6  746.72  5073.0  749.58  5077.1  748.17  5080.4  753.69  5081.2  747.08
  5084.8  755.77  5101.0  765.51  5102.4  762.23  5102.8  747.94  5109.4  770.76
  5153.7  794.94  5258.7  839.31  5271.9  857.91  5280.9  849.12  5327.0  865.67
#Mann=3,-1,0
  4568.0    0.15       0  4967.3    0.05       0  5032.7    0.15       0
Bank Sta=4967.3,5032.7
XS Rating Curve= 0
Exp/Cntr=0.3,0.1

Type RM Length L Ch R = 1,51907,407,407,407
BEGIN DESCRIPTION:
Chauga River 104.0
END DESCRIPTION:
XS GIS Cut Line= 4
      1354070.35      1045838.96      1353682.21      1045524.57
      1353570.49      1045446.21      1353358.83      1045425.81
#Sta/Elev= 30
  4500.5  825.42  4544.4  822.12  4600.3  812.71  4717.7  784.87  4770.4  774.83
  4842.2  756.75  4850.5  753.48  4875.3  750.83  4895.1  745.23  4932.7  744.57
  4940.3  742.66  4961.6  731.16  4961.8  733.57  4967.3  731.16  4967.8  730.16
  5032.2  730.16  5032.7  731.16  5047.6  731.16  5066.3  739.70  5067.6  738.62
  5071.2  738.71  5099.0  741.26  5130.4  744.62  5145.4  747.35  5160.4  751.90
  5167.5  752.98  5206.9  767.18  5269.8  781.69  5303.1  792.70  5349.1  803.80
#Mann=3,-1,0
  4500.5    0.15       0  4967.3    0.05       0  5032.7    0.15       0
Bank Sta=4967.3,5032.7
XS Rating Curve= 0
Exp/Cntr=0.3,0.1

Type RM Length L Ch R = 1,51500,500,500,500
BEGIN DESCRIPTION:
Chauga River 103.0
END DESCRIPTION:
XS GIS Cut Line= 3
      1353751.53      1045023.41      1353512.59      1045226.67
      1353328.25      1045372.74
#Sta/Elev= 30
  4686.3  784.75  4738.1  784.37  4773.9  782.45  4816.9  772.00  4859.2  756.16
  4874.8  753.40  4881.7  749.18  4897.2  741.84  4898.0  737.22  4907.9  736.62
  4919.3  733.89  4922.9  732.11  4938.1  735.94  4955.2  735.88  4966.9  733.56
  4967.3  728.50  4967.8  727.50  5032.2  727.50  5032.7  728.50  5035.1  728.50
  5036.3  730.10  5049.8  740.30  5060.3  745.56  5091.1  748.79  5103.3  751.54
  5136.1  767.11  5164.0  778.41  5174.3  783.52  5219.7  800.78  5235.2  807.79
#Mann=3,-1,0
  4686.3    0.15       0  4967.3    0.05       0  5032.7    0.15       0
Bank Sta=4967.3,5032.7
XS Rating Curve= 0
Exp/Cntr=0.3,0.1

Type RM Length L Ch R = 1,51000,500,500,500
BEGIN DESCRIPTION:
Chauga River 102.0
END DESCRIPTION:
XS GIS Cut Line= 3
      1353557.78      1044770.90      1353193.73      1044845.41
      1352726.37      1045020.83
#Sta/Elev= 30
  4628.4  783.14  4672.9  777.20  4734.8  758.92  4738.1  754.95  4746.1  755.88
  4845.0  745.86  4916.6  742.94  4939.8  739.10  4952.3  730.96  4953.4  728.50
  4967.3  728.50  4967.8  727.50  5032.7  728.50  5035.8  728.50  5046.3  736.90
  5055.2  741.38  5061.1  741.69  5063.9  745.30  5097.6  757.29  5100.7  759.81
  5107.9  758.36  5132.2  763.48  5133.5  762.23  5145.3  764.38  5223.2  785.85
  5293.0  813.38  5326.5  829.90  5371.0  848.86  5435.7  872.33  5499.2  891.63
#Mann=3,-1,0
  4628.4    0.15       0  4967.3    0.05       0  5032.7    0.15       0
Bank Sta=4967.3,5032.7
XS Rating Curve= 0
Exp/Cntr=0.3,0.1

Type RM Length L Ch R = 1,50500,500,500,500
BEGIN DESCRIPTION:
Chauga River 101.0
END DESCRIPTION:
XS GIS Cut Line= 3
      1353590.90      1044620.20      1353315.15      1044425.26
      1352922.77      1044176.48
#Sta/Elev= 30
  4662.3  767.75  4684.2  774.91  4724.5  775.59  4738.8  770.39  4753.9  767.68
  4797.1  762.32  4871.2  748.40  4925.5  741.75  4947.8  737.05  4958.3  728.50
  4962.7  731.36  4967.3  728.50  4967.8  727.50  5032.7  728.50  5033.3  731.27
  5051.0  739.66  5061.9  741.60  5080.3  753.94  5100.1  757.40  5117.5  763.38
  5128.1  763.32  5152.4  769.14  5229.1  771.69  5268.3  775.07  5271.7  777.62
  5283.7  780.35  5299.0  778.41  5307.5  779.11  5309.2  781.98  5464.6  793.49
#Mann=3,-1,0
  4662.3    0.15       0  4967.3    0.05       0  5032.7    0.15       0
Bank Sta=4967.3,5032.7
XS Rating Curve= 0
Exp/Cntr=0.3,0.1

Type RM Length L Ch R = 1,50000,500,500,500
BEGIN DESCRIPTION:
Chauga River 100.0
END DESCRIPTION:
XS GIS Cut Line= 3
      1353797.46      1044388.11      1353725.96      1044148.76
      1353672.51      1043838.83
#Sta/Elev= 30
  4750.2  784.65  4782.5  780.65  4810.4  774.94  4889.6  746.58  4942.1  735.58
  4953.9  731.22  4956.2  729.93  4956.5  728.50  4967.3  727.21  4967.8  726.21
  5032.2  726.21  5032.7  727.21  5045.0  735.86  5048.4  728.50  5048.8  732.38
  5058.9  739.30  5072.6  752.52  5075.0  744.14  5075.2  741.58  5075.6  750.23
  5077.4  754.00  5079.0  755.05  5080.5  748.79  5081.2  736.14  5085.3  754.83
  5136.2  768.76  5249.1  789.72  5274.8  792.35  5292.1  791.05  5314.5  792.29
#Mann=3,-1,0
  4750.2    0.15       0  4967.3    0.05       0  5032.7    0.15       0
Bank Sta=4967.3,5032.7
XS Rating Curve= 0
Exp/Cntr=0.3,0.1

Type RM Length L Ch R = 1,49500,500,500,500
BEGIN DESCRIPTION:
Chauga River 99.0
END DESCRIPTION:
XS GIS Cut Line= 3
      1353981.06      1044404.98      1354192.85      1044145.94
      1354389.11      1043917.86
#Sta/Elev= 30
  4665.4  801.20  4678.4  801.29  4687.7  797.90  4722.4  791.92  4746.8  783.87
  4880.7  747.70  4911.0  742.64  4967.3  728.39  4967.8  727.39  5032.7  728.39
  5053.3  728.50  5070.2  735.94  5082.2  750.65  5083.0  750.03  5085.3  740.61
  5085.8  755.88  5086.7  755.95  5089.7  738.78  5089.8  752.45  5096.5  765.25
  5109.2  769.75  5117.8  778.81  5123.6  782.02  5151.7  787.06  5169.4  785.68
  5175.7  787.19  5193.4  792.69  5232.2  810.52  5266.8  820.78  5300.9  828.26
#Mann=3,-1,0
  4665.4    0.15       0  4967.3    0.05       0  5032.7    0.15       0
Bank Sta=4967.3,5032.7
XS Rating Curve= 0
Exp/Cntr=0.3,0.1

Type RM Length L Ch R = 1,49000,500,500,500
BEGIN DESCRIPTION:
Chauga River 98.0
END DESCRIPTION:
XS GIS Cut Line= 3
      1354845.58      1044440.62      1354624.96      1044145.59
      1354457.97      1043917.85
#Sta/Elev= 30
  4631.6  801.17  4661.4  792.74  4703.3  776.20  4741.0  774.42  4741.4  773.80
  4741.6  765.79  4753.4  776.31  4767.4  771.39  4834.0  765.86  4887.5  730.85
  4923.9  720.93  4967.2  719.20  4967.7  718.20  5032.8  719.20  5067.3  727.01
  5072.1  732.26  5085.9  740.31  5096.6  740.96  5104.3  744.97  5118.8  762.32
  5144.8  776.88  5171.2  779.74  5201.3  793.39  5248.2  810.40  5254.4  793.44
  5259.8  791.65  5259.9  788.83  5260.0  796.05  5265.2  816.48  5282.4  822.11
#Mann=3,-1,0
  4631.6    0.15       0  4967.2    0.05       0  5032.8    0.15       0
Bank Sta=4967.2,5032.8
XS Rating Curve= 0
Exp/Cntr=0.3,0.1

Type RM Length L Ch R = 1,48500,676,676,676
BEGIN DESCRIPTION:
Chauga River 97.0
END DESCRIPTION:
XS GIS Cut Line= 3
      1355057.27      1043673.55      1354764.06      1043690.45
      1354491.12      1043757.71
#Sta/Elev= 30
  4706.3  800.91  4717.8  798.40  4747.0  798.37  4753.3  797.15  4754.4  795.51
  4789.4  790.79  4800.0  785.53  4835.7  773.63  4872.9  767.71  4889.9  762.37
  4912.0  745.21  4935.8  731.38  4940.3  723.87  4943.8  726.44  4959.2  718.99
  4966.4  710.31  4966.8  712.12  4967.2  710.31  4967.7  709.31  5032.8  710.31
  5036.0  715.61  5041.3  717.15  5063.5  721.70  5068.4  720.90  5072.7  723.85
  5081.6  723.14  5106.0  741.10  5152.1  768.06  5249.4  813.81  5281.1  832.64
#Mann=3,-1,0
  4706.3    0.15       0  4967.2    0.05       0  5032.8    0.15       0
Bank Sta=4967.2,5032.8
XS Rating Curve= 0
Exp/Cntr=0.3,0.1

Type RM Length L Ch R = 1,47824,324,324,324
BEGIN DESCRIPTION:
Chauga River 96.0
END DESCRIPTION:
XS GIS Cut Line= 3
      1354859.46      1042814.78      1354643.73      1043087.33
      1354338.33      1043386.34
#Sta/Elev= 30
  4652.4  755.10  4694.8  757.34  4732.2  761.98  4759.0  762.31  4781.5  766.11
  4830.0  762.72  4857.6  763.01  4865.6  756.11  4871.0  758.41  4881.3  755.78
  4911.9  753.78  4930.2  740.13  4933.5  740.17  4937.2  735.56  4938.0  728.05
  4941.6  733.09  4943.9  720.41  4945.3  717.32  4964.2  715.79  4966.1  707.82
  4966.6  706.82  5033.9  707.82  5064.9  710.41  5089.1  716.72  5095.9  714.71
  5159.8  719.79  5222.3  748.56  5268.3  763.37  5380.5  779.59  5427.4  788.49
#Mann=3,-1,0
  4652.4    0.15       0  4966.1    0.05       0  5033.9    0.15       0
Bank Sta=4966.1,5033.9
XS Rating Curve= 0
Exp/Cntr=0.3,0.1

Type RM Length L Ch R = 1,47500,500,500,500
BEGIN DESCRIPTION:
Chauga River 95.0
END DESCRIPTION:
XS GIS Cut Line= 3
      1354533.44      1042738.14      1354340.06      1042979.41
      1354125.43      1043202.26
#Sta/Elev= 30
  4690.8  800.11  4751.8  791.78  4753.5  796.70  4761.8  789.73  4818.9  774.58
  4866.1  757.31  4881.9  755.41  4889.8  751.28  4911.0  731.71  4916.7  736.10
  4924.9  715.50  4925.0  720.51  4929.0  725.13  4935.7  720.10  4940.7  713.00
  4943.0  706.28  4943.8  710.45  4966.1  706.28  4966.6  705.28  5033.9  706.28
  5045.6  706.28  5064.6  714.90  5077.7  724.17  5083.6  724.92  5099.4  734.66
  5120.7  750.79  5136.8  759.71  5178.5  776.39  5246.7  795.31  5309.4  805.33
#Mann=3,-1,0
  4690.8    0.15       0  4966.1    0.05       0  5033.9    0.15       0
Bank Sta=4966.1,5033.9
XS Rating Curve= 0
Exp/Cntr=0.3,0.1

Type RM Length L Ch R = 1,47000,500,500,500
BEGIN DESCRIPTION:
Chauga River 94.0
END DESCRIPTION:
XS GIS Cut Line= 3
      1354268.24      1042266.32      1354014.80      1042609.22
      1353829.61      1042880.91
#Sta/Elev= 30
  4573.6  864.13  4681.7  842.34  4754.5  821.27  4769.7  819.28  4779.3  824.12
  4803.1  807.13  4828.6  799.37  4839.4  792.85  4854.2  778.39  4870.4  776.25
  4887.3  764.60  4903.1  746.09  4916.6  722.85  4917.8  708.47  4919.0  720.45
  4920.8  723.97  4923.7  718.04  4932.0  711.27  4932.4  731.28  4932.9  722.03
  4939.2  702.37  4943.2  699.07  4947.7  701.52  4966.1  698.90  4966.6  697.90
  5033.9  698.90  5105.7  715.04  5137.4  717.35  5197.8  728.90  5328.8  772.90
#Mann=3,-1,0
  4573.6    0.15       0  4966.1    0.05       0  5033.9    0.15       0
Bank Sta=4966.1,5033.9
XS Rating Curve= 0
Exp/Cntr=0.3,0.1

Type RM Length L Ch R = 1,46500,500,500,500
BEGIN DESCRIPTION:
Chauga River 93.0
END DESCRIPTION:
XS GIS Cut Line= 3
      1353521.02      1042159.25      1353546.61      1042493.27
      1353572.03      1042942.15
#Sta/Elev= 30
  4665.0  783.42  4766.9  746.63  4769.3  755.64  4770.5  784.05  4771.5  764.25
  4771.6  744.86  4846.2  712.30  4850.9  711.47  4852.8  715.23  4856.2  704.94
  4860.8  708.97  4869.9  706.64  4871.9  703.71  4878.9  699.73  4890.8  700.46
  4929.3  695.24  4963.8  695.37  4966.1  692.84  4966.6  691.84  5033.4  691.84
  5033.9  692.84  5106.8  707.56  5167.6  733.77  5208.4  748.92  5243.8  755.93
  5254.3  759.74  5296.8  768.00  5394.8  780.66  5423.4  786.77  5449.6  795.21
#Mann=3,-1,0
  4665.0    0.15       0  4966.1    0.05       0  5033.9    0.15       0
Bank Sta=4966.1,5033.9
XS Rating Curve= 0
Exp/Cntr=0.3,0.1

Type RM Length L Ch R = 1,46000,500,500,500
BEGIN DESCRIPTION:
Chauga River 92.0
END DESCRIPTION:
XS GIS Cut Line= 3
      1353222.63      1042200.04      1353055.55      1042551.66
      1352883.46      1042891.14
#Sta/Elev= 30
  4610.7  768.94  4696.4  754.32  4698.2  760.27  4698.4  757.24  4704.9  750.79
  4728.2  743.34  4773.1  707.04  4786.4  703.37  4787.3  727.96  4788.4  704.72
  4788.8  702.91  4869.8  699.43  4938.3  703.72  4962.8  699.22  4963.3  698.61
  4963.8  692.26  4966.1  689.94  4966.6  688.94  5033.9  689.94  5048.1  695.92
  5053.1  712.22  5057.7  711.38  5081.9  731.12  5146.8  767.59  5163.3  773.30
  5199.8  778.57  5226.4  774.04  5263.7  787.96  5303.6  796.01  5380.6  797.16
#Mann=3,-1,0
  4610.7    0.15       0  4966.1    0.05       0  5033.9    0.15       0
Bank Sta=4966.1,5033.9
XS Rating Curve= 0
Exp/Cntr=0.3,0.1

Type RM Length L Ch R = 1,45500,539,539,539
BEGIN DESCRIPTION:
Chauga River 91.0
END DESCRIPTION:
XS GIS Cut Line= 3
      1352929.34      1042046.78      1352669.89      1042242.51
      1352335.13      1042633.34
#Sta/Elev= 30
  4675.0  753.93  4706.2  756.15  4729.3  753.64  4808.7  736.78  4842.4  726.20
  4855.5  719.33  4859.8  721.01  4897.7  718.83  4912.8  713.96  4926.6  706.26
  4943.6  699.78  4960.0  688.20  4966.1  687.80  4966.6  686.80  5033.4  686.80
  5033.9  687.80  5040.2  700.04  5041.1  698.15  5073.0  701.56  5126.1  702.80
  5135.2  705.03  5140.1  703.16  5142.1  706.14  5165.4  714.28  5199.2  731.38
  5241.8  746.41  5253.1  747.05  5308.7  743.70  5461.9  746.33  5514.6  748.95
#Mann=3,-1,0
  4675.0    0.15       0  4966.1    0.05       0  5033.9    0.15       0
Bank Sta=4966.1,5033.9
XS Rating Curve= 0
Exp/Cntr=0.3,0.1

Type RM Length L Ch R = 1,44961,461,461,461
BEGIN DESCRIPTION:
Chauga River 90.0
END DESCRIPTION:
XS GIS Cut Line= 3
      1352845.25      1041960.04      1352193.15      1042015.97
      1351554.75      1041993.20
#Sta/Elev= 30
  4345.5  738.36  4441.9  733.71  4478.5  725.98  4646.9  711.80  4786.5  710.59
  4904.0  702.28  4916.5  698.98  4931.1  687.63  4966.1  687.57  4966.6  686.57
  5033.9  687.57  5048.0  687.57  5048.2  691.11  5052.3  695.19  5072.3  702.98
  5159.0  708.04  5160.3  716.71  5162.6  722.42  5167.8  716.86  5175.0  728.63
  5180.7  727.19  5182.4  735.00  5192.1  717.78  5245.8  740.72  5389.2  731.33
  5500.1  748.00  5519.5  755.98  5527.0  772.66  5530.0  761.43  5638.8  780.24
#Mann=3,-1,0
  4345.5    0.15       0  4966.1    0.05       0  5033.9    0.15       0
Bank Sta=4966.1,5033.9
XS Rating Curve= 0
Exp/Cntr=0.3,0.1

Type RM Length L Ch R = 1,44500,500,500,500
BEGIN DESCRIPTION:
Chauga River 89.0
END DESCRIPTION:
XS GIS Cut Line= 3
      1352829.45      1041806.21      1352481.46      1041678.43
      1352146.49      1041581.55
#Sta/Elev= 30
  4629.3  747.99  4668.7  756.50  4686.5  752.95  4710.0  754.17  4774.1  744.44
  4819.7  735.37  4909.6  705.68  4946.0  702.11  4959.5  697.36  4965.4  692.63
  4966.1  687.03  4966.6  686.03  5033.9  687.03  5062.8  701.85  5069.4  716.91
  5070.0  721.01  5076.4  708.77  5086.8  707.00  5087.6  703.89  5087.7  710.41
  5088.4  716.34  5107.2  741.99  5183.5  775.36  5184.6  783.85  5186.1  780.48
  5186.4  777.09  5190.5  778.12  5241.9  802.60  5291.8  821.46  5348.7  835.32
#Mann=3,-1,0
  4629.3    0.15       0  4966.1    0.05       0  5033.9    0.15       0
Bank Sta=4966.1,5033.9
XS Rating Curve= 0
Exp/Cntr=0.3,0.1

Type RM Length L Ch R = 1,44000,540,540,540
BEGIN DESCRIPTION:
Chauga River 88.0
END DESCRIPTION:
XS GIS Cut Line= 3
      1353197.91      1041419.77      1352773.93      1041274.74
      1352532.92      1041222.07
#Sta/Elev= 30
  4551.9  787.02  4591.9  784.65  4678.6  782.66  4723.7  778.71  4776.2  771.35
  4810.1  761.04  4867.5  739.53  4874.1  741.10  4892.2  735.99  4915.0  717.28
  4930.2  714.55  4950.0  701.31  4957.9  700.09  4959.5  696.90  4963.3  696.19
  4966.1  686.04  4966.6  685.04  5033.4  685.04  5033.9  686.04  5041.1  691.18
  5046.7  697.42  5047.8  700.08  5049.0  698.62  5082.9  704.11  5104.8  705.39
  5117.9  709.39  5140.1  710.23  5144.7  712.19  5160.7  713.80  5246.7  745.40
#Mann=3,-1,0
  4551.9    0.15       0  4966.1    0.05       0  5033.9    0.15       0
Bank Sta=4966.1,5033.9
XS Rating Curve= 0
Exp/Cntr=0.3,0.1

Type RM Length L Ch R = 1,43460,460,460,460
BEGIN DESCRIPTION:
Chauga River 87.0
END DESCRIPTION:
XS GIS Cut Line= 3
      1353181.29      1040623.76      1352970.15      1040793.48
      1352600.16      1041072.81
#Sta/Elev= 30
  4729.1  727.71  4776.5  723.18  4807.6  717.25  4845.3  712.86  4871.8  707.99
  4897.2  706.26  4911.3  703.18  4929.3  701.22  4940.5  695.69  4944.8  694.33
  4945.4  696.27  4959.7  690.25  4966.0  685.32  4966.5  684.32  5033.5  684.32
  5034.0  685.32  5035.6  697.69  5035.9  697.95  5058.2  700.87  5072.4  704.39
  5074.2  706.12  5080.2  703.95  5118.4  707.46  5267.1  706.67  5310.8  708.87
  5363.9  714.70  5419.7  729.49  5443.1  738.25  5455.4  738.11  5463.6  739.07
#Mann=3,-1,0
  4729.1    0.15       0  4966.0    0.05       0  5034.0    0.15       0
Bank Sta=4966,5034
XS Rating Curve= 0
Exp/Cntr=0.3,0.1

Type RM Length L Ch R = 1,43000,394,394,394
BEGIN DESCRIPTION:
Chauga River 86.0
END DESCRIPTION:
XS GIS Cut Line= 4
      1352578.55      1040455.62      1352612.05      1040608.80
      1352645.80      1040902.30      1352561.76      1041091.98
#Sta/Elev= 30
  4843.2  744.88  4895.8  745.30  4898.9  748.40  4900.9  753.02  4902.1  751.73
  4903.7  757.35  4906.3  747.43  4913.0  739.58  4916.8  738.53  4925.0  729.83
  4942.8  715.94  4956.6  696.48  4958.1  698.74  4964.7  717.14  4966.0  683.61
  4966.5  682.61  5034.0  683.61  5041.4  688.77  5046.0  688.41  5054.6  696.49
  5062.7  697.99  5068.2  702.10  5077.6  703.32  5135.9  701.97  5191.6  709.94
  5257.5  714.29  5262.6  712.94  5272.7  716.57  5341.0  725.66  5502.9  740.51
#Mann=3,-1,0
  4843.2    0.15       0  4966.0    0.05       0  5034.0    0.15       0
Bank Sta=4966,5034
XS Rating Curve= 0
Exp/Cntr=0.3,0.1

Type RM Length L Ch R = 1,42606,223,223,223
BEGIN DESCRIPTION:
Chauga River 85.0
END DESCRIPTION:
XS GIS Cut Line= 4
      1352483.14      1040525.43      1352316.21      1040671.11
      1352269.17      1040794.60      1352165.52      1041243.28
#Sta/Elev= 30
  4646.3  738.60  4666.7  738.14  4686.8  735.30  4716.8  727.80  4754.7  723.00
  4766.5  718.76  4775.6  706.40  4794.3  702.63  4810.2  700.68  4863.8  699.91
  4882.7  697.57  4930.6  698.58  4955.5  684.88  4966.0  683.24  4966.5  682.24
  5034.0  683.24  5039.8  685.92  5054.9  696.61  5069.5  700.89  5085.2  700.55
  5117.1  707.00  5125.5  707.47  5137.6  704.35  5323.2  704.35  5335.1  710.28
  5349.3  709.53  5364.1  711.97  5379.6  719.88  5432.5  734.00  5460.5  744.26
#Mann=3,-1,0
  4646.3    0.15       0  4966.0    0.05       0  5034.0    0.15       0
Bank Sta=4966,5034
XS Rating Curve= 0
Exp/Cntr=0.3,0.1

Type RM Length L Ch R = 1,42383,383,383,383
BEGIN DESCRIPTION:
Chauga River 84.5
END DESCRIPTION:
XS GIS Cut Line= 4
      1352455.89      1040513.23      1352261.57      1040634.69
      1352152.83      1040649.53      1351848.69      1040671.11
#Sta/Elev= 30
  4661.1  730.20  4683.8  727.43  4725.2  717.20  4781.1  707.04  4855.9  699.98
  4903.1  697.91  4942.4  698.86  4951.8  693.78  4956.3  689.85  4959.2  684.95
  4959.4  683.62  4962.9  685.60  4965.8  682.85  4966.3  681.85  5033.7  681.85
  5034.2  682.85  5036.0  690.43  5043.0  698.01  5048.2  695.38  5062.0  698.91
  5089.9  714.42  5108.0  722.04  5116.5  728.06  5118.0  726.18  5144.9  736.03
  5196.5  750.48  5225.6  757.15  5243.4  763.31  5285.8  763.13  5304.9  761.52
#Mann=3,-1,0
  4661.1    0.15       0  4965.8    0.05       0  5034.2    0.15       0
Bank Sta=4965.8,5034.2
XS Rating Curve= 0
Exp/Cntr=0.3,0.1

Type RM Length L Ch R = 1,42000,500,500,500
BEGIN DESCRIPTION:
Chauga River 84.0
END DESCRIPTION:
XS GIS Cut Line= 3
      1352667.71      1040386.29      1352271.51      1040289.31
      1351849.92      1040161.62
#Sta/Elev= 30
  4592.1  763.85  4713.7  727.66  4767.6  714.66  4814.5  710.51  4885.1  709.15
  4896.2  706.66  4902.3  701.20  4916.7  704.30  4921.9  697.36  4930.2  702.90
  4952.4  695.47  4965.6  687.04  4965.8  681.73  4966.3  680.73  5034.2  681.73
  5041.4  695.95  5044.8  695.58  5049.4  700.15  5066.5  704.99  5078.0  711.43
  5118.0  743.27  5150.9  763.73  5189.5  784.00  5219.2  796.77  5261.1  805.25
  5292.7  805.61  5332.6  800.89  5410.7  782.81  5426.6  782.40  5440.5  778.22
#Mann=3,-1,0
  4592.1    0.15       0  4965.8    0.05       0  5034.2    0.15       0
Bank Sta=4965.8,5034.2
XS Rating Curve= 0
Exp/Cntr=0.3,0.1

Type RM Length L Ch R = 1,41500,500,500,500
BEGIN DESCRIPTION:
Chauga River 83.0
END DESCRIPTION:
XS GIS Cut Line= 3
      1352964.30      1040134.67      1352450.08      1039823.19
      1351939.75      1039523.53
#Sta/Elev= 30
  4398.8  776.06  4502.7  755.04  4511.0  750.95  4550.6  740.98  4568.9  739.98
  4579.0  734.65  4602.5  729.92  4628.3  729.70  4640.5  724.74  4687.7  714.76
  4717.6  711.23  4907.0  703.75  4910.8  700.76  4932.3  696.09  4958.2  696.12
  4965.7  692.31  4965.8  679.99  4966.3  678.99  5034.2  679.99  5050.2  692.80
  5099.4  714.44  5117.0  716.51  5118.5  719.40  5123.3  716.88  5145.5  718.35
  5190.9  725.61  5289.4  747.50  5375.5  756.91  5499.7  758.88  5591.8  764.08
#Mann=3,-1,0
  4398.8    0.15       0  4965.8    0.05       0  5034.2    0.15       0
Bank Sta=4965.8,5034.2
XS Rating Curve= 0
Exp/Cntr=0.3,0.1

Type RM Length L Ch R = 1,41000,500,500,500
BEGIN DESCRIPTION:
Chauga River 82.0
END DESCRIPTION:
XS GIS Cut Line= 3
      1353224.97      1039724.98      1352766.78      1039436.41
      1352274.99      1039275.00
#Sta/Elev= 30
  4458.5  758.41  4585.1  742.54  4726.8  714.41  4797.9  706.73  4870.9  704.29
  4925.0  705.05  4941.4  698.05  4948.0  697.83  4951.3  693.27  4961.4  688.72
  4965.8  680.54  4966.3  679.54  5034.2  680.54  5037.1  687.47  5041.2  689.12
  5046.0  693.99  5079.3  697.21  5127.9  723.59  5153.2  733.02  5176.8  738.76
  5187.5  737.65  5200.9  739.33  5231.1  736.85  5270.2  740.47  5276.6  739.51
  5312.4  745.17  5331.2  751.68  5380.5  761.36  5423.4  766.92  5517.6  774.70
#Mann=3,-1,0
  4458.5    0.15       0  4965.8    0.05       0  5034.2    0.15       0
Bank Sta=4965.8,5034.2
XS Rating Curve= 0
Exp/Cntr=0.3,0.1

Type RM Length L Ch R = 1,40500,500,500,500
BEGIN DESCRIPTION:
Chauga River 81.0
END DESCRIPTION:
XS GIS Cut Line= 3
      1353575.02      1039275.01      1353096.99      1039062.11
      1352730.67      1038953.79
#Sta/Elev= 30
  4476.7  797.74  4595.2  777.46  4599.1  780.51  4604.8  776.28  4667.3  764.73
  4700.3  754.60  4772.1  724.79  4811.7  711.77  4834.2  705.93  4875.5  699.57
  4946.0  694.96  4965.0  687.00  4965.8  679.50  4966.3  678.50  5034.2  679.50
  5038.2  681.15  5039.9  685.28  5050.1  688.49  5051.0  691.54  5051.3  695.38
  5054.6  692.51  5091.1  701.76  5152.5  726.02  5168.2  736.57  5189.4  738.13
  5197.7  742.35  5228.4  748.26  5288.2  752.52  5329.5  749.97  5382.0  743.31
#Mann=3,-1,0
  4476.7    0.15       0  4965.8    0.05       0  5034.2    0.15       0
Bank Sta=4965.8,5034.2
XS Rating Curve= 0
Exp/Cntr=0.3,0.1

Type RM Length L Ch R = 1,40000,500,500,500
BEGIN DESCRIPTION:
Chauga River 80.0
END DESCRIPTION:
XS GIS Cut Line= 3
      1353539.41      1038333.71      1353083.11      1038675.48
      1352586.86      1038962.75
#Sta/Elev= 30
  4429.9  801.71  4454.3  798.98  4477.4  786.74  4514.1  784.40  4519.4  777.81
  4519.8  782.75  4526.7  779.69  4577.8  780.34  4610.3  772.73  4652.9  769.05
  4735.1  778.30  4812.7  774.12  4864.8  756.36  4893.2  754.54  4916.7  744.56
  4927.4  731.47  4945.4  716.94  4953.4  719.05  4964.3  695.42  4964.8  699.36
  4965.8  679.57  4966.3  678.57  5034.2  679.57  5057.5  692.38  5111.2  696.46
  5169.9  707.34  5292.2  736.10  5351.4  740.12  5445.1  734.73  5573.4  747.10
#Mann=3,-1,0
  4429.9    0.15       0  4965.8    0.05       0  5034.2    0.15       0
Bank Sta=4965.8,5034.2
XS Rating Curve= 0
Exp/Cntr=0.3,0.1

Type RM Length L Ch R = 1,39500,500,500,500
BEGIN DESCRIPTION:
Chauga River 79.0
END DESCRIPTION:
XS GIS Cut Line= 3
      1352974.98      1038075.02      1352637.75      1038449.98
      1352274.97      1038825.03
#Sta/Elev= 30
  4495.7  760.65  4531.2  760.99  4542.6  763.95  4549.7  770.67  4645.6  764.27
  4667.1  775.31  4713.9  756.49  4755.2  749.10  4777.0  739.32  4779.0  742.45
  4782.0  762.09  4782.1  753.04  4783.2  749.62  4784.6  737.65  4861.0  720.97
  4892.5  706.53  4939.7  694.28  4943.7  696.05  4944.2  701.37  4952.2  693.32
  4957.8  680.07  4965.8  677.76  4966.3  676.76  5034.2  677.76  5038.6  691.57
  5057.0  697.14  5185.0  713.92  5275.8  742.40  5428.2  768.70  5521.8  775.66
#Mann=3,-1,0
  4495.7    0.15       0  4965.8    0.05       0  5034.2    0.15       0
Bank Sta=4965.8,5034.2
XS Rating Curve= 0
Exp/Cntr=0.3,0.1

Type RM Length L Ch R = 1,39000,500,500,500
BEGIN DESCRIPTION:
Chauga River 78.0
END DESCRIPTION:
XS GIS Cut Line= 3
      1352625.03      1037874.98      1352220.35      1038177.24
      1351774.99      1038825.01
#Sta/Elev= 30
  4494.9  771.62  4544.9  778.82  4568.5  779.15  4577.1  772.57  4582.1  766.72
  4583.1  762.64  4584.5  765.78  4616.1  765.29  4638.1  771.34  4661.3  769.54
  4707.0  753.52  4724.2  752.82  4845.2  705.78  4905.4  695.91  4952.6  692.63
  4963.1  686.46  4965.8  677.60  4966.3  676.60  5034.2  677.60  5038.5  693.13
  5071.6  698.81  5119.8  695.84  5151.9  700.74  5214.4  703.80  5276.7  714.38
  5364.2  719.45  5498.6  752.34  5612.8  784.17  5689.8  812.61  5786.1  834.23
#Mann=3,-1,0
  4494.9    0.15       0  4965.8    0.05       0  5034.2    0.15       0
Bank Sta=4965.8,5034.2
XS Rating Curve= 0
Exp/Cntr=0.3,0.1

Type RM Length L Ch R = 1,38500,500,500,500
BEGIN DESCRIPTION:
Chauga River 77.0
END DESCRIPTION:
XS GIS Cut Line= 3
      1352002.69      1037544.61      1351810.70      1037892.21
      1351526.38      1038578.12
#Sta/Elev= 30
  4602.9  765.62  4695.2  749.60  4707.3  751.44  4745.6  740.93  4794.4  723.65
  4804.6  717.88  4857.6  704.53  4936.7  699.16  4955.5  691.37  4957.2  686.48
  4963.1  684.49  4965.8  676.56  4966.3  675.56  5034.2  676.56  5038.5  689.73
  5048.4  693.60  5065.1  692.11  5156.9  697.80  5210.8  698.04  5211.5  695.48
  5212.6  697.53  5242.4  703.03  5322.2  728.87  5365.6  737.57  5405.0  740.63
  5494.3  735.97  5600.4  747.67  5681.4  760.92  5721.7  754.72  5742.5  758.67
#Mann=3,-1,0
  4602.9    0.15       0  4965.8    0.05       0  5034.2    0.15       0
Bank Sta=4965.8,5034.2
XS Rating Curve= 0
Exp/Cntr=0.3,0.1

Type RM Length L Ch R = 1,38000,500,500,500
BEGIN DESCRIPTION:
Chauga River 76.0
END DESCRIPTION:
XS GIS Cut Line= 3
      1351575.00      1037325.01      1351335.23      1037768.20
      1351125.01      1038424.98
#Sta/Elev= 30
  4496.1  761.46  4549.6  766.84  4576.6  766.09  4600.3  761.24  4701.2  724.88
  4772.7  703.64  4811.3  696.93  4811.8  698.72  4854.6  696.66  4904.4  697.63
  4924.8  693.60  4941.2  693.94  4965.1  684.52  4965.8  676.41  4966.3  675.41
  5034.2  676.41  5040.4  686.75  5042.2  687.79  5056.7  689.50  5085.1  702.06
  5108.4  707.53  5152.5  713.16  5173.2  712.29  5265.8  716.78  5309.8  724.58
  5356.5  741.87  5406.8  757.35  5414.4  761.84  5642.3  817.57  5689.6  827.13
#Mann=3,-1,0
  4496.1    0.15       0  4965.8    0.05       0  5034.2    0.15       0
Bank Sta=4965.8,5034.2
XS Rating Curve= 0
Exp/Cntr=0.3,0.1

Type RM Length L Ch R = 1,37500,500,500,500
BEGIN DESCRIPTION:
Chauga River 75.0
END DESCRIPTION:
XS GIS Cut Line= 3
      1351175.00      1037174.99      1350869.67      1037592.57
      1350525.02      1037974.98
#Sta/Elev= 30
  4482.7  762.21  4531.9  761.69  4563.6  756.43  4684.4  742.61  4689.9  739.88
  4798.8  716.75  4855.8  701.27  4883.1  697.87  4930.9  697.54  4949.5  689.51
  4956.5  689.02  4962.0  683.12  4965.8  675.61  4966.3  674.61  5034.2  675.61
  5035.8  686.78  5050.7  688.70  5050.9  690.38  5067.7  696.79  5106.4  716.48
  5110.4  721.08  5123.6  725.18  5161.3  742.95  5287.8  774.31  5350.8  784.94
  5394.6  804.04  5400.9  810.03  5408.2  814.18  5466.8  842.83  5514.8  861.35
#Mann=3,-1,0
  4482.7    0.15       0  4965.8    0.05       0  5034.2    0.15       0
Bank Sta=4965.8,5034.2
XS Rating Curve= 0
Exp/Cntr=0.3,0.1

Type RM Length L Ch R = 1,37000,660,660,660
BEGIN DESCRIPTION:
Chauga River 74.0
END DESCRIPTION:
XS GIS Cut Line= 3
      1350873.07      1037038.28      1350525.75      1037232.84
      1350079.15      1037469.21
#Sta/Elev= 30
  4601.9  740.83  4643.2  734.76  4690.5  732.80  4730.5  722.15  4773.0  708.47
  4821.3  699.73  4833.3  700.64  4866.4  697.67  4938.3  697.59  4944.4  694.47
  4949.7  693.99  4958.0  688.18  4965.8  674.78  4966.3  673.78  5034.2  674.78
  5035.3  680.48  5048.4  689.04  5076.8  695.17  5128.0  717.34  5154.9  727.50
  5180.5  734.45  5213.7  737.49  5317.6  736.69  5339.2  734.73  5379.6  724.00
  5411.4  724.95  5448.7  720.38  5462.9  727.39  5499.3  733.19  5505.3  737.11
#Mann=3,-1,0
  4601.9    0.15       0  4965.8    0.05       0  5034.2    0.15       0
Bank Sta=4965.8,5034.2
XS Rating Curve= 0
Exp/Cntr=0.3,0.1

Type RM Length L Ch R = 1,36340,443,443,443
BEGIN DESCRIPTION:
Chauga River 73.0
END DESCRIPTION:
XS GIS Cut Line= 3
      1350772.86      1036968.48      1350109.32      1036761.41
      1349755.95      1036580.70
#Sta/Elev= 30
  4304.9  730.26  4465.7  715.35  4507.3  703.04  4540.4  704.42  4554.1  697.52
  4555.3  704.55  4584.2  696.59  4656.2  698.22  4675.1  693.21  4790.8  689.05
  4829.1  684.31  4884.3  686.12  4933.6  692.39  4944.6  690.69  4957.6  683.45
  4965.8  672.90  4966.3  671.90  5034.2  672.90  5034.7  681.92  5049.0  687.67
  5058.5  697.24  5088.6  703.63  5107.0  714.82  5121.9  718.76  5150.5  712.14
  5161.7  705.64  5342.0  705.35  5386.1  709.81  5388.3  707.10  5396.9  710.53
#Mann=3,-1,0
  4304.9    0.15       0  4965.8    0.05       0  5034.2    0.15       0
Bank Sta=4965.8,5034.2
XS Rating Curve= 0
Exp/Cntr=0.3,0.1

Type RM Length L Ch R = 1,35897,397,397,397
BEGIN DESCRIPTION:
Chauga River 72.0
END DESCRIPTION:
XS GIS Cut Line= 3
      1350775.57      1036925.54      1350482.81      1036533.86
      1350165.57      1036346.76
#Sta/Elev= 30
  4511.0  735.33  4519.4  736.35  4540.6  730.87  4590.9  724.61  4614.7  716.07
  4709.8  710.57  4752.2  710.10  4781.6  707.96  4830.7  700.68  4908.2  695.51
  4948.0  689.84  4956.6  687.23  4965.3  683.52  4965.8  672.36  4966.3  671.36
  5034.2  672.36  5037.8  674.59  5040.9  680.22  5045.4  684.26  5065.4  691.96
  5121.6  697.28  5195.5  700.61  5214.2  702.70  5238.3  707.89  5275.0  709.01
  5285.7  711.50  5304.9  711.19  5356.0  714.20  5366.0  716.07  5368.3  715.03
#Mann=3,-1,0
  4511.0    0.15       0  4965.8    0.05       0  5034.2    0.15       0
Bank Sta=4965.8,5034.2
XS Rating Curve= 0
Exp/Cntr=0.3,0.1
